HEC-RAS study 04072003_Bear_Creek.prj: Bear Creek

--- 04072003_Bear_Creek.g01 (geometry) --- (continued)

Type RM Length L Ch R = 1 ,24913.0,502.3,502.3,502.3
BEGIN DESCRIPTION:
Cross Section Bear Creek 32.0
END DESCRIPTION:
#Sta/Elev= 30
  3822.9   70.55  3842.9   68.83  3937.9   63.84  4072.9   59.54  4252.9   57.98
  4261.3   57.55  4272.9   56.95  4337.9   55.48  4407.9   53.29  4441.8   53.32
  4841.8   51.26 4973.95   51.79 4976.35   50.32 4978.15    49.5 4981.65   48.72
 4998.55    49.9 5017.55   47.58 5023.15   50.23 5026.05   51.18  5106.8   53.28
  5206.8   59.17  5372.7   60.72  5437.7   60.92  5457.7   62.09  5492.7   61.11
  5517.7    61.2  5526.9   61.87  5542.7   63.01  5584.7    63.7  5602.9      64
#Mann= 6 , 1 , 0
 3822.90     0.1       0  4261.3    0.14       0 4973.95   0.045       0
 5026.05    0.14       0  5526.9     0.1       0  5584.7     0.2       0
Bank Sta=4973.95,5026.05
Exp/Cntr=0.5,0.3

Type RM Length L Ch R = 1 ,24410.7,46.2,46.2,46.2
BEGIN DESCRIPTION:
Upstream Section of Bridge/Culvert/Weir
END DESCRIPTION:
#Sta/Elev= 30
  4009.1   71.66  4084.1   64.76  4129.1   62.73  4274.1   59.99  4586.3   57.21
  4687.1   53.31  4742.1   53.44  4768.6   54.63  4870.7   52.52  4926.2   52.53
  4969.3    56.6  4981.4   50.81  4990.8   50.65  4998.5   47.58  5011.6   50.61
  5015.4   48.76  5034.4   46.44  5042.9   50.04    5054   50.36  5067.9   55.45
  5160.2    53.4  5212.7   55.59  5377.5   54.28  5407.5   55.98  5452.5   55.54
  5537.5   60.73  5623.7   61.16  5782.3   61.08  6077.8   63.38  6127.8   66.02
#Mann= 7 , 1 , 0
 4009.10     0.2       0  4009.1     0.1       0  4586.3    0.14       0
  4990.8   0.045       0  5042.9    0.14       0  5623.7     0.1       0
  6077.8     0.2       0
#XS Ineff= 2 , 0
       0    4965    58.4    5065       0    57.8
Bank Sta=4990.80,5042.90
Exp/Cntr=0.5,0.3

Type RM Length L Ch R = 3 ,24387.6,,,
BEGIN DESCRIPTION:
MAYS STORE RD
Structure ID: L_BEACR2
END DESCRIPTION:
Bridge Culvert--1,0,-1,-1, 0
Deck Dist Width WeirC Skew NumUp NumDn MinLoCord MaxHiCord MaxSubmerge Is_Ogee
10,26.2,2.6,, 57, 57,,,0.95,0,1,1,,
  4009.1  4014.1  4034.1  4054.1  4084.1  4119.1  4129.1  4164.5  4189.5  4259.5
  4274.1  4292.5  4372.5  4497.1  4592.1  4662.1  4672.1  4687.1  4727.1  4732.1
  4742.1  4768.6  4822.1  4870.7  4926.2  4969.3  4974.9 4975.01  4975.1 4975.33
 4975.44 5055.19  5055.3 5055.69  5055.8 5055.91  5067.9  5106.7  5160.2  5212.7
  5270.3  5360.8  5377.5  5407.5  5412.5  5427.5  5452.5  5537.5  5667.3  5692.3
  5700.8  5722.3  5782.3  6007.3  6012.3  6077.8  6127.8
   71.64   70.77   69.25   67.11   64.74   63.31   62.71    62.9   62.64   60.73
   60.13   59.76   59.01   58.85   58.72   58.54   58.52   58.48   58.52   58.53
   58.55   58.61   58.71   58.68   58.64   58.53   58.51   58.36   58.23   57.91
   60.91    61.5    61.5    60.8    60.8    57.8   57.92   58.29   58.38   58.46
   58.47    58.1   58.26   58.56   58.61   58.75      59   60.72   61.36    61.5
    61.6   61.14   61.06   62.31   62.98   63.36      66
   71.64   70.77   69.25   67.11   64.74   63.31   62.71   62.04   61.57   60.25
   59.97   59.75   58.81   57.35   57.18   54.14   54.08   53.29   54.43   54.32
   53.42   54.61      54    52.5   52.51   56.58    53.9   53.85   56.13   55.81
   55.81    56.4   50.82   50.96      51   51.04   55.43   54.28   53.38   55.57
   54.63   54.32   54.26   55.96   56.01   55.09   55.52   60.71   61.35   61.42
   61.34   61.14   61.06   62.31   62.98   63.36      66
  4009.1  4014.1  4034.1  4054.1  4084.1  4119.1  4129.1  4164.5  4189.5  4259.5
  4274.1  4292.5  4372.5  4497.1  4592.1  4662.1  4672.1  4687.1  4727.1  4732.1
  4742.1  4768.6  4822.1  4870.7  4926.2  4969.3  4974.9 4975.01  4975.1 4975.33
 4975.44 5055.19  5055.3 5055.69  5055.8 5055.91  5067.9  5106.7  5160.2  5212.7
  5270.3  5360.8  5377.5  5407.5  5412.5  5427.5  5452.5  5537.5  5667.3  5692.3
  5700.8  5722.3  5782.3  6007.3  6012.3  6077.8  6127.8
   71.64   70.77   69.25   67.11   64.74   63.31   62.71    62.9   62.64   60.73
   60.13   59.76   59.01   58.85   58.72   58.54   58.52   58.48   58.52   58.53
   58.55   58.61   58.71   58.68   58.64   58.53   58.51   58.36   58.23   57.91
   60.91    61.5    61.5    60.8    60.8    57.8   57.92   58.29   58.38   58.46
   58.47    58.1   58.26   58.56   58.61   58.75      59   60.72   61.36    61.5
    61.6   61.14   61.06   62.31   62.98   63.36      66
   71.54   70.67   69.15   67.01   64.64   63.21   62.61   61.94   61.47   60.15
   59.87   59.65   58.71   57.25   57.08   54.04   53.98   53.19   54.33   54.22
   53.32   54.51    53.9    52.4   52.41   56.48    53.8   53.75   56.03   55.71
   55.71    56.3   50.72   50.86    50.9   50.94   55.33   54.18   53.28   55.47
   54.53   54.22   54.16   55.86   55.91   54.99   55.42   60.61   61.25   61.32
   61.24   61.04   60.96   62.21   62.88   63.26    65.9
Pier Skew, UpSta & Num, DnSta & Num=,4995.0, 2 ,4995.0, 2 , 0 , 0 , 0 ,,
       1       1
   47.23   56.95
       1       1
   47.13   56.85
Pier Skew, UpSta & Num, DnSta & Num=,5015.4, 2 ,5015.4, 2 , 0 , 0 , 0 ,,
       1       1
   47.68    57.1
       1       1
   47.58      57
Pier Skew, UpSta & Num, DnSta & Num=,5034.4, 2 ,5034.4, 2 , 0 , 0 , 0 ,,
       1       1
   45.49   57.25
       1       1
   45.39   57.15
Abutment Skew #Up #Dn=, 2 , 2
 4974.90 4981.50
   56.13   50.79
 4974.90 4981.50
   56.03   50.69
Abutment Skew #Up #Dn=, 2 , 2
 5054.10 5055.39
   50.38   56.40
 5054.10 5055.39
   50.28   56.30
BR Coef= 1 , 1 , 0 ,1.25, 0 ,,,0.8,0,2,0,
Wspro=,,,, 1 ,,,, 0 ,,,, 0 ,,,,-1 ,-1 ,-1 , 0 , 0 , 0 , 0 , 0
BC Design=,, 0 ,, 0 ,,,,,,
BR U #Sta/Elev= 92
  4009.1   71.64  4014.1   70.77  4034.1   69.25  4054.1   67.11  4084.1   64.74
  4119.1   63.31  4129.1   62.71  4164.5   62.04  4189.5   61.57  4194.5   61.47
  4259.5   60.25  4272.5      60  4274.1   59.97  4292.5   59.75  4372.5   58.81
  4497.1   57.35  4586.3   57.19  4589.5   57.18  4592.1   57.18  4662.1   54.14
  4672.1   54.08  4687.1   53.29  4698.6   53.62  4727.1   54.43  4732.1   54.32
  4742.1   53.42  4761.4   54.29  4768.6   54.61  4817.5   54.05  4822.1      54
  4868.5   52.57  4870.7    52.5  4923.2   52.51  4926.2   52.51  4969.3   56.58
  4974.9    53.9 4975.01   53.85  4975.1    53.8 4975.33   53.69 4975.44   53.64
 4975.55   53.59  4981.4   50.79  4981.5   50.79  4990.8   50.63  4993.2   49.16
    4995   48.34  4998.5   47.56  5006.8   49.13  5011.6   50.59  5014.6    49.3
  5015.4   48.74  5031.3   46.86  5034.4   46.42    5040   49.07  5042.9   50.02
    5054   50.34  5054.1   50.38 5055.19   50.78  5055.3   50.82  5055.4   50.85
 5055.69   50.96  5055.8      51 5055.91   51.04  5067.9   55.43  5106.7   54.28
  5108.4   54.25  5160.2   53.38  5160.9   53.41  5212.7   55.57  5213.1   55.56
  5270.3   54.63  5274.7   54.61  5360.8   54.32  5377.5   54.26  5407.5   55.96
  5412.5   56.01  5427.5   55.09  5452.5   55.52  5537.5   60.71  5607.5   61.06
  5623.7   61.14  5635.8    61.2  5667.3   61.35  5692.3   61.42  5700.8   61.34
  5722.3   61.14  5782.3   61.06  6007.3   62.31  6012.3   62.98  6077.7   63.36
  6077.8   63.36  6127.8      66
BR U #Mann= 7
 4009.10     0.2  4009.1     0.1  4586.3    0.14  4990.8   0.045  5042.9    0.14
  5623.7     0.1  6077.8     0.2
BR U Banks=4990.80,5042.90
BR D #Sta/Elev= 92
  4009.1   71.54  4014.1   70.67  4034.1   69.15  4054.1   67.01  4084.1   64.64
  4119.1   63.21  4129.1   62.61  4164.5   61.94  4189.5   61.47  4194.5   61.37
  4259.5   60.15  4272.5    59.9  4274.1   59.87  4292.5   59.65  4372.5   58.71
  4497.1   57.25  4586.3   57.09  4589.5   57.08  4592.1   57.08  4662.1   54.04
  4672.1   53.98  4687.1   53.19  4698.6   53.52  4727.1   54.33  4732.1   54.22
  4742.1   53.32  4761.4   54.19  4768.6   54.51  4817.5   53.95  4822.1    53.9
  4868.5   52.47  4870.7    52.4  4923.2   52.41  4926.2   52.41  4969.3   56.48
  4974.9    53.8 4975.01   53.75  4975.1    53.7 4975.33   53.59 4975.44   53.54
 4975.55   53.49  4981.4   50.69  4981.5   50.69  4990.8   50.53  4993.2   49.06
    4995   48.24  4998.5   47.46  5006.8   49.03  5011.6   50.49  5014.6    49.2
  5015.4   48.64  5031.3   46.76  5034.4   46.32    5040   48.97  5042.9   49.92
    5054   50.24  5054.1   50.28 5055.19   50.68  5055.3   50.72  5055.4   50.75
 5055.69   50.86  5055.8    50.9 5055.91   50.94  5067.9   55.33  5106.7   54.18
  5108.4   54.15  5160.2   53.28  5160.9   53.31  5212.7   55.47  5213.1   55.46
  5270.3   54.53  5274.7   54.51  5360.8   54.22  5377.5   54.16  5407.5   55.86
  5412.5   55.91  5427.5   54.99  5452.5   55.42  5537.5   60.61  5607.5   60.96
  5623.7   61.04  5635.8    61.1  5667.3   61.25  5692.3   61.32  5700.8   61.24
  5722.3   61.04  5782.3   60.96  6007.3   62.21  6012.3   62.88  6077.7   63.26
  6077.8   63.26  6127.8    65.9
BR D #Mann= 7
 4009.10     0.2  4009.1     0.1  4586.3    0.14  4990.8   0.045  5042.9    0.14
  5623.7     0.1  6077.8     0.2
BR D Banks=4990.80,5042.90

Type RM Length L Ch R = 1 ,24364.5,969.5,969.5,969.5
BEGIN DESCRIPTION:
Downstream Section of Bridge/Culvert/Weir
END DESCRIPTION:
#Sta/Elev= 30
  4009.1   71.53  4084.1   64.63  4129.1    62.6  4274.1   59.86  4586.3   57.08
  4687.1   53.18  4742.1   53.31  4768.6    54.5  4870.7   52.39  4926.2    52.4
  4969.3   56.47  4981.4   50.68  4990.8   50.52  4998.5   47.45  5011.6   50.48
  5015.4   48.63  5034.4   46.31  5042.9   49.91    5054   50.23  5067.9   55.32
  5160.2   53.27  5212.7   55.46  5377.5   54.15  5407.5   55.85  5452.5   55.41
  5537.5    60.6  5623.7   61.03  5782.3   60.95  6077.8   63.25  6127.8   65.89
#Mann= 7 , 1 , 0
 4009.10     0.2       0  4009.1     0.1       0  4586.3    0.14       0
  4990.8   0.045       0  5042.9    0.14       0  5623.7     0.1       0
  6077.8     0.2       0
#XS Ineff= 2 , 0
       0    4965    57.4    5065       0    57.4
Bank Sta=4990.80,5042.90
Exp/Cntr=0.5,0.3

Type RM Length L Ch R = 1 ,23395.0,806,806,806
BEGIN DESCRIPTION:
Cross Section Bear Creek 31.0
END DESCRIPTION:
#Sta/Elev= 30
  3598.5   63.99  3608.5   63.42  3703.5   62.17  3723.5      61  3753.5   60.85
  3773.5   59.48  3817.3   58.89  4020.1   58.62  4318.5   57.54  4343.5   56.91
  4618.5   57.09  4663.5   55.71  4863.5   52.02  4908.5   51.81 4973.95   49.71
 4978.15   47.42 4981.65   46.64 4998.55   47.82 5017.55    45.5 5026.05    49.1
  5212.3   51.73  5222.3   52.45  5312.3   52.72  5422.3   54.47  5532.3   54.08
  5572.3   55.23  5627.3   59.79  5643.2   60.26  5712.3   60.24  5782.3   61.69
#Mann= 7 , 1 , 0
 3598.50     0.2       0  3598.5    0.15       0  3817.3     0.1       0
  4020.1    0.15       0 4973.95   0.045       0 5026.05    0.15       0
  5643.2     0.1       0
Bank Sta=4973.95,5026.05
Exp/Cntr=0.3,0.1

Type RM Length L Ch R = 1 ,22589.0,423,423,423
BEGIN DESCRIPTION:
Cross Section Bear Creek 30.0
END DESCRIPTION:
#Sta/Elev= 30
  3614.4   65.11  3624.4   63.74  3644.4   62.31  3654.4   61.12  3784.4   58.56
  3934.4    57.7  4089.4   54.52  4164.4   54.62  4219.4   54.41  4429.4   55.55
  4546.2   53.49  4599.4   52.46  4689.4   52.47  4976.5   51.76  4979.6    48.2
  4981.6   44.82  5002.6   47.08    5016   47.22  5019.7   48.21  5023.5   50.89
  5087.9   51.11  5157.9   50.62  5602.9   53.22  5685.1   57.63  5695.1   57.73
  5785.1   61.86  5793.9   61.82  5865.1    61.5  6260.1   61.01  6437.3   62.16
#Mann= 7 , 1 , 0
 3614.40     0.2       0  3614.4     0.1       0  4546.2    0.15       0
  4976.5   0.045       0  5023.5    0.15       0  5793.9     0.1       0
  6437.3     0.2       0
Bank Sta=4976.50,5023.50
Exp/Cntr=0.3,0.1

Type RM Length L Ch R = 1 ,22166.0,739,739,739
BEGIN DESCRIPTION:
Cross Section CCX_L68
Located At: CCX_L68 CNTRL
END DESCRIPTION:
#Sta/Elev= 30
  3525.1   64.23  3600.1   61.33  3625.1   58.68  3720.1   57.76  4110.1   58.85
  4260.1   55.65  4370.1   54.51  4425.1   55.33  4467.3   53.72  4540.1   50.96
  4600.1   51.56  4680.1   50.84  4725.1   51.59  4802.6   50.81  4952.9    52.2
  4976.8   51.41  4979.9   47.85  4981.9   44.47  5002.9   46.73  5016.3   46.87
    5020   47.86  5023.8   51.54  5069.9   50.01  5352.6   53.05  5387.6   51.37
  5497.6   51.96  5712.6   56.13  5938.4   55.58  6048.4   56.18  6098.4   62.48
#Mann= 5 , 1 , 0
 3525.10     0.2       0  3525.1     0.1       0  4467.3    0.15       0
  4976.8   0.045       0  5023.8    0.15       0
Bank Sta=4976.80,5023.80
Exp/Cntr=0.3,0.1

Type RM Length L Ch R = 1 ,21427.0,628,628,628
BEGIN DESCRIPTION:
Cross Section Bear Creek 29.0
END DESCRIPTION:
#Sta/Elev= 28
  3685.7   60.68  3780.7   57.92  4180.7   57.15  4345.7   53.73  4499.1   53.51
  4505.7    53.5  4650.7   53.97  4680.7   52.45  4690.7   51.66  4755.7   50.03
  4830.7   50.46  4885.7   50.27  4976.5   50.05  4979.6   46.49  4981.6   43.11
  5002.6   45.37    5016   45.51  5019.7    46.5  5023.5   49.18  5071.9    49.6
  5216.9   49.63  5226.9   49.87  5251.9   50.63  5286.9   56.06  5301.9    56.9
  5321.9   57.39  5381.9   61.15  5451.9    61.4
#Mann= 5 , 1 , 0
 3685.70     0.2       0  3685.7     0.1       0  4499.1    0.15       0
  4976.5   0.045       0  5023.5    0.15       0
Bank Sta=4976.50,5023.50
Exp/Cntr=0.3,0.1

Type RM Length L Ch R = 1 ,20799.0,451,451,451
BEGIN DESCRIPTION:
Cross Section Bear Creek 28.0
END DESCRIPTION:
#Sta/Elev= 30
  3248.1   61.05  3513.1   56.64  3903.1   58.02  4143.1   54.63  4208.1   54.47
  4388.1   55.79  4508.1   55.06  4540.4   54.06  4558.1   53.51  4648.1   53.07
  4658.1   53.54  4703.1   53.53  4743.1   52.91  4803.1   49.94 4980.55   50.19
 4985.75   43.35 5008.05   45.69 5011.25    46.7 5017.35   47.16 5019.45   49.34
  5167.9   49.36  5227.9   51.59  5302.9   51.52  5377.9   53.82  5462.9   52.23
  5489.9   53.27  5499.9   54.24  5579.9   57.36  5624.1   56.93  5833.3   60.05
#Mann= 7 , 1 , 0
 3248.10     0.2       0  3248.1     0.1       0  4540.4    0.15       0
 4980.55   0.045       0 5019.45    0.15       0  5624.1     0.1       0
  5833.3     0.2       0
Bank Sta=4980.55,5019.45
Exp/Cntr=0.3,0.1

Type RM Length L Ch R = 1 ,20348.0,579,579,579
BEGIN DESCRIPTION:
Cross Section Bear Creek 27.0
END DESCRIPTION:
#Sta/Elev= 30
  3134.3   60.42  3229.3    58.7  3869.3   58.41  4019.3   54.01  4114.3   54.71
  4254.3   54.45  4442.6   54.83  4516.5   53.14  4582.6   51.69  4592.6   52.53
  4627.6   52.48  4645.3   51.82  4750.3   50.86  4785.3   48.06 4980.55   47.42
 4983.05   45.92 4985.75   42.58 5008.05   44.92 5011.25   45.93 5017.35   46.39
 5019.45   48.57  5034.1   47.82  5054.1   49.24  5119.1   49.21  5179.1   52.02
  5239.1   52.26  5249.1   53.07  5418.8   54.52  5689.1   60.13  5719.1   60.21
#Mann= 6 , 1 , 0
 3134.30     0.2       0  3134.3     0.1       0  4516.5    0.15       0
 4980.55   0.045       0 5019.45    0.15       0  5418.8     0.1       0
Bank Sta=4980.55,5019.45
Exp/Cntr=0.3,0.1

Type RM Length L Ch R = 1 ,19769.0,712,712,712
BEGIN DESCRIPTION:
Cross Section Bear Creek 26.0
END DESCRIPTION:
#Sta/Elev= 30
  2970.3   59.96  3230.3   58.06  3480.3   59.07  3750.3   58.65  4200.3   59.32
  4311.7   59.38  4461.7   58.55  4481.7   58.93  4508.2   57.71  4531.7    56.2
  4546.7   56.06  4611.7   50.74  4661.7   50.19  4721.7   51.39  4841.7   48.77
 4980.55   48.39 4985.75   42.55 5017.35   46.36 5019.45   49.54  5138.5   49.25
  5308.5   50.87  5318.5   51.89  5478.5    53.4  5483.5    52.9  5587.8   52.41
  5597.8   53.48  5647.8   54.65  5772.8   59.27  5782.8   60.07  5822.8   60.87
#Mann= 5 , 1 , 0
 2970.30      10       0  4200.3     0.1       0  4508.2    0.15       0
 4980.55   0.045       0 5019.45    0.15       0
Bank Sta=4980.55,5019.45
Exp/Cntr=0.3,0.1

Type RM Length L Ch R = 1 ,19057.0,621,621,621
BEGIN DESCRIPTION:
Cross Section Bear Creek 25.0
END DESCRIPTION:
#Sta/Elev= 30
  2693.9   61.08  2858.9   57.59  3273.9   58.11  3408.9   56.59  3418.9   57.61
  3643.9   56.73  3863.9   57.72  4078.9   57.24  4199.9   58.55  4320.3   56.49
  4516.9   51.85  4656.9   50.99  4711.9   48.24  4761.9   49.49  4781.9   48.25
  4821.9   49.51  4956.9   50.14 4980.55   48.83 4985.75   41.99 5017.35    45.8
 5019.45   47.98  5087.9   48.47  5117.9   46.81  5272.9   53.22  5357.9   52.72
    5500   57.16  5582.9   57.48  5617.9   56.03  5817.9   53.36  5922.9   61.27
#Mann= 6 , 1 , 0
 2693.90      10       0  4199.9     0.1       0  4320.3    0.15       0
 4980.55   0.045       0 5019.45    0.15       0    5500      10       0
Bank Sta=4980.55,5019.45
Exp/Cntr=0.3,0.1

Type RM Length L Ch R = 1 ,18436.0,623,623,623
BEGIN DESCRIPTION:
Cross Section CCX_L23
Located At: CCX_L23 CTRL
END DESCRIPTION:
#Sta/Elev= 30
    4021   58.66    4226   57.34    4353    54.6    4476   52.36    4521   53.31
  4579.5   51.94  4604.5   50.33  4629.5   50.22  4644.5   49.26  4689.5   50.21
  4769.5   49.32  4794.5   47.95  4874.5   49.05  4921.3   47.81  4983.4      48
  4988.6   41.16  5020.2   44.97  5022.3   48.15    5041   47.75  5065.4   49.22
  5170.6   48.06  5240.8   54.58  5280.8    56.5  5475.8   57.12  5625.8   55.72
  5710.8    56.6  5900.8   55.39  5940.8   58.15    5966   58.26  6314.8    58.4
#Mann= 7 , 1 , 0
 4021.00     0.2       0    4021     0.1       0    4353    0.15       0
  4983.4   0.045       0  5022.3    0.15       0    5966     0.1       0
  6314.8     0.2       0
Bank Sta=4983.40,5022.30
Exp/Cntr=0.3,0.1

Type RM Length L Ch R = 1 ,17813.0,513,513,513
BEGIN DESCRIPTION:
Cross Section Bear Creek 24.0
END DESCRIPTION:
#Sta/Elev= 30
  3920.6    58.7  4270.6   57.05  4410.6   52.66  4440.6   50.79  4480.6    50.6
  4606.5   52.58  4625.6    53.1  4710.6   52.48  4880.6   47.69  4945.6   47.84
  4975.6   45.01 4980.55   47.38 4985.75   40.54 5017.35   44.35 5019.45   46.53
  5224.5   47.14  5359.5   54.57  5399.6   54.17  5444.5   53.73  5489.5   51.46
  5641.3   53.94  5666.3   53.24  5696.3      54  6026.3   54.59  6066.3    53.3
  6146.3    53.9  6196.3   57.17  6211.3   57.46  6676.3   56.85  6811.7   58.43
#Mann= 5 , 1 , 0
 3920.60     0.1       0  4606.5    0.15       0 4980.55   0.045       0
 5019.45    0.15       0  5399.6      10       0
Bank Sta=4980.55,5019.45
Exp/Cntr=0.3,0.1

Type RM Length L Ch R = 1 ,17300.0,445,445,445
BEGIN DESCRIPTION:
Cross Section Bear Creek 23.0
END DESCRIPTION:
#Sta/Elev= 30
  3817.7   58.82  3827.7   58.22  3932.7   57.84  4027.7   56.48  4222.7   56.81
  4297.7   55.93  4315.8   54.96  4352.7   52.98  4417.7    51.4  4447.7   51.74
  4482.7   50.01  4532.7   50.15  4627.7   48.85  4716.5    46.9  4736.5   47.09
  4791.5   46.24  4811.5   47.53 4980.55   47.18 4985.75   40.34 5017.35   44.15
 5019.45   47.33  5209.8   51.02  5389.8   49.01  5709.8   52.95  5734.8   52.27
  5944.1   54.26  6103.5   57.13  6374.1   56.25  6654.1   57.08  6767.4   58.11
#Mann= 7 , 1 , 0
 3817.70     0.2       0  3817.7     0.1       0  4315.8    0.15       0
 4980.55   0.045       0 5019.45    0.15       0  6103.5     0.1       0
  6767.4     0.2       0
Bank Sta=4980.55,5019.45
Exp/Cntr=0.3,0.1

Type RM Length L Ch R = 1 ,16855.0,406,406,406
BEGIN DESCRIPTION:
Cross Section Bear Creek 22.0
END DESCRIPTION:
#Sta/Elev= 30
  4249.9   58.21  4339.9   55.41  4390.9   53.06  4409.9   52.19  4449.9   48.31
  4459.9   47.98  4484.9   47.68  4509.9   48.51  4579.9   48.12  4809.9   46.61
  4924.9   44.73 4980.55      45 4983.05    43.5 4985.75   40.16 5017.35   43.97
 5019.45   47.15  5279.6   49.04  5364.6   50.31  5409.6   50.24  5429.6   49.18
  5464.6   49.62  5489.6    51.3  5499.6   51.09  5594.6   55.34  5725.2    55.4
  5962.8   56.81  6110.8   55.99  6321.8   56.99  6361.8   57.98  6724.9   58.01
#Mann= 8 , 1 , 0
 4249.90     0.1       0  4390.9    0.15       0 4980.55   0.045       0
 5019.45    0.15       0  5725.2     0.1       0  5962.8    0.15       0
  6110.8     0.1       0  6724.9     0.2       0
Bank Sta=4980.55,5019.45
Exp/Cntr=0.3,0.1

Type RM Length L Ch R = 1 ,16449.0,700,700,700
BEGIN DESCRIPTION:
Cross Section Bear Creek 21.0
END DESCRIPTION:
#Sta/Elev= 30
  3967.3    57.9  4132.3   56.59  4182.3   56.49  4391.4   51.44  4407.3   51.06
  4462.3   50.53  4487.3   49.16  4497.3   47.73  4582.3   47.68  4667.3    48.1
  4702.3   47.27  4797.3   46.53  4957.3   46.76  4977.2   47.08  4987.1   42.67
  4989.4    41.9  5003.1   40.15  5014.6   39.19  5017.3   42.85  5022.8   47.91
  5052.9   48.76  5357.9   50.35  5372.9   51.44  5472.9   51.92  5627.9   52.21
  5657.9   55.26  5662.9   55.58  5672.6   55.79  5687.9   56.12  6244.2   57.19
#Mann= 5 , 1 , 0
 3967.30     0.1       0  4391.4    0.15       0  4977.2   0.045       0
  5022.8    0.15       0  5672.6     0.1       0
Bank Sta=4977.20,5022.80
Exp/Cntr=0.3,0.1

Type RM Length L Ch R = 1 ,15749.0,707,707,707
BEGIN DESCRIPTION:
Cross Section Bear Creek 20.0
END DESCRIPTION:
#Sta/Elev= 30
  4092.6   56.41  4382.6   54.24  4417.6      53  4437.6   52.76  4447.6   52.16
  4462.6   51.93  4472.6   51.24  4488.1   51.12  4572.6   50.41  4602.6   50.74
  4782.6   50.06  4812.6   49.69  4917.6   49.48  4977.2   46.81  4987.1    42.4
  4989.4   41.63  5003.1   39.88  5014.6   38.92  5017.3   42.58  5022.8   47.64
  5197.3   48.06  5232.3   48.68  5502.3    50.8  5542.3   50.81  5687.3   51.76
  5777.3   55.77  5794.4   55.89  5907.3   57.11  6443.8   58.12  6443.9   58.12
#Mann= 7 , 1 , 0
 4092.60     0.2       0  4092.6     0.1       0  4488.1    0.15       0
  4977.2   0.045       0  5022.8    0.15       0  5794.4     0.1       0
  6443.8     0.2       0
Bank Sta=4977.20,5022.80
Exp/Cntr=0.3,0.1

Type RM Length L Ch R = 1 ,15042.0,467,467,467
BEGIN DESCRIPTION:
Cross Section CCX_L67
Located At: CCX_L67 CTRL
END DESCRIPTION:
#Sta/Elev= 30
  3698.6   56.16  3918.6   55.33  4008.6   53.15  4133.6   51.37  4223.6   51.05
  4333.6   49.85  4497.2   49.51    4513   49.04  4597.2   48.58  4632.2   47.19
  4925.9   46.96  4950.3   45.18    4975   46.07  4987.2   40.89  5012.4   38.18
  5015.1   41.84  5020.6    46.9  5067.5   46.36  5192.5   46.25  5257.5   51.39
  5362.7   52.78  5577.5   53.72  5617.5   54.54  5702.5   54.32  5787.5   53.08
  5972.5   53.66  6042.5   55.83  6057.5   56.72  6121.4   57.87  6427.2   58.14
#Mann= 7 , 1 , 0
 3698.60     0.2       0  3698.6     0.1       0    4513    0.15       0
    4975   0.045       0  5020.6    0.15       0  5362.7     0.1       0
  6427.2     0.2       0
Bank Sta=4975.00,5020.60
Exp/Cntr=0.3,0.1

Type RM Length L Ch R = 1 ,14575.0,692,692,692
BEGIN DESCRIPTION:
Cross Section Bear Creek 19.0
END DESCRIPTION:
#Sta/Elev= 30
  4042.5    56.5  4157.5   55.55  4236.8   55.58  4262.5   54.89  4267.5   53.66
  4307.5   51.66  4437.5   51.45  4467.5   50.77  4522.5   47.63  4672.5   44.85
  4732.5   45.35  4966.7   42.37  4969.8   40.29  4996.4   40.03    5006   39.25
  5013.3   37.66  5020.1   37.67  5030.3   39.36  5031.9    40.5  5033.3    43.2
  5082.9   44.63  5182.9    45.2  5257.9   46.65  5272.9   48.18  5347.9    50.8
  5467.9    53.2  5492.9   54.41    5533   54.22  5737.9   55.56  5905.2   57.37
#Mann= 6 , 1 , 0
 4042.50     0.1       0  4236.8    0.15       0  4966.7   0.045       0
  5033.3    0.15       0    5533     0.1       0  5905.2     0.2       0
Bank Sta=4966.70,5033.30
Exp/Cntr=0.3,0.1

Type RM Length L Ch R = 1 ,13883.0,744,744,744
BEGIN DESCRIPTION:
Cross Section Bear Creek 18.0
END DESCRIPTION:
#Sta/Elev= 30
  4402.2   56.45  4462.2   55.29  4472.2   55.58  4663.3   51.75  4682.2   52.02
  4742.2   47.48  4792.2    44.8  4862.2   42.11  4966.7   42.22  4969.8   40.14
  4996.4   39.88    5006    39.1  5013.3   37.51  5020.1   37.52  5030.3   39.21
  5031.9   40.35  5033.3   43.05  5047.3   44.28  5162.3   43.46  5237.3   44.15
  5272.3   44.99  5372.3   45.08  5462.3   46.35  5517.3   48.85    5638   50.38
  5652.3   50.73  5662.3   50.58  5795.9   54.76  6085.9   54.95  6200.9    56.6
#Mann= 6 , 1 , 0
 4402.20     0.2       0  4402.2     0.1       0  4663.3    0.15       0
  4966.7   0.045       0  5033.3    0.15       0    5638     0.1       0
Bank Sta=4966.70,5033.30
Exp/Cntr=0.3,0.1

Type RM Length L Ch R = 1 ,13139.0,805,805,805
BEGIN DESCRIPTION:
Cross Section Bear Creek 17.0
END DESCRIPTION:
#Sta/Elev= 30
  4376.7   54.95  4505.2   54.75  4591.7   54.17  4746.7    51.1  4806.7   50.86
  4811.7   50.47  4866.7   42.22  4966.7   42.01  4969.8   39.93  4996.4   39.67
    5006   38.89  5013.3    37.3  5020.1   37.31  5030.3      39  5031.9   40.14
  5033.3   42.84  5054.7   42.93  5094.7   45.28  5249.7    44.4  5539.7   46.92
  5629.7   49.47  5649.7   48.73  5694.7   48.13  5729.7   48.18  5963.6   50.47
  6100.1   52.37  6137.1   53.23  6242.1   53.61  6253.8   54.07  6464.8   56.38
#Mann= 9 , 1 , 0
 4376.70     0.2       0  4376.7     0.1       0  4505.2    0.15       0
  4966.7   0.045       0  5033.3    0.15       0  5963.6     0.1       0
  6100.1    0.15       0  6253.8     0.1       0  6464.8     0.2       0
Bank Sta=4966.70,5033.30
Exp/Cntr=0.3,0.1

Type RM Length L Ch R = 1 ,12334.0,756.65,756.65,756.65
BEGIN DESCRIPTION:
Cross Section Bear Creek 16.0
END DESCRIPTION:
#Sta/Elev= 30
  4178.1   55.24  4228.1    54.2  4348.1   53.74  4363.1   51.97  4378.1    51.5
  4453.1   50.62  4538.1   49.91  4658.1   50.53  4813.1   45.02  4966.7   42.43
  4969.8   39.35  4996.4   39.09    5006   38.31  5013.3   36.72  5020.1   36.73
  5030.3   38.42  5031.9   39.56  5033.3   42.26  5096.7    43.7  5361.7    44.6
  5371.7   46.23  5401.7    48.8    5419   49.04  5471.7   49.32  5491.7   50.34
  5541.7   51.13  5577.1   50.95  5842.5    50.8  5906.7    54.7  5967.6   55.17
#Mann= 8 , 1 , 0
 4178.10     0.2       0  4178.1    0.15       0  4966.7   0.045       0
  5033.3    0.15       0    5419     0.1       0  5577.1    0.15       0
  5842.5     0.1       0  5967.6     0.2       0
Bank Sta=4966.70,5033.30
Exp/Cntr=0.5,0.3

Type RM Length L Ch R = 1 ,11577.4,40.7,40.7,40.7
BEGIN DESCRIPTION:
Upstream Section of Bridge/Culvert/Weir
END DESCRIPTION:
#Sta/Elev= 30
  4196.5   54.73  4321.5   52.59  4496.5   45.53  4601.9   43.76  4848.1    43.8
  4897.2   42.87  4945.3   43.63  4962.2   43.31  4965.9   41.83    4969   38.75
  4995.6   38.49  5012.5   36.12  5019.3   36.13  5029.5   37.82  5031.1   38.96
  5032.5   41.66  5050.6   47.43  5107.3   48.19  5132.4    47.4  5222.9   45.83
  5296.9   46.95  5451.1   47.83  5672.7   50.43  5682.7   49.61  5697.7   50.56
  5762.7   50.23  5800.8   51.41  5900.8   52.39  5935.8   51.93  6115.8   54.35
#Mann= 6 , 1 , 0
 4196.50    0.15       0  4965.9   0.045       0  5032.5    0.15       0
  5132.4    0.14       0  5296.9    0.15       0  5451.1    0.14       0
#XS Ineff= 2 , 0
       0    4935    48.7    5067       0    48.4
Bank Sta=4965.90,5032.50
Exp/Cntr=0.5,0.3

Type RM Length L Ch R = 3 ,11557.0,,,
BEGIN DESCRIPTION:
BEAR CREEK RD
Structure ID: L_BEACR1
END DESCRIPTION:
Bridge Culvert--1,0,-1,-1, 0
Deck Dist Width WeirC Skew NumUp NumDn MinLoCord MaxHiCord MaxSubmerge Is_Ogee
10,20.7,2.6,, 47, 47,,,0.95,0,1,1,,
  4196.5  4231.5  4286.5  4301.5  4321.5  4395.8  4496.5  4601.9  4661.7  4741.7
  4795.9  4848.1  4897.2  4922.9 4944.61 4944.72 4944.83  4944.9  4945.1  4945.2
  4945.3 5048.19  5048.3 5056.99  5057.1  5057.2  5107.3  5167.9  5222.9    5275
  5312.7  5337.6  5387.7  5427.6  5497.6  5672.7  5677.7  5682.7  5697.7  5762.7
  5775.8  5800.8  5890.8  5900.8  5935.8  6105.8  6115.8
   54.72   54.07   52.78   52.84   52.59   49.58   48.37   48.26   48.19   48.68
   48.85   48.78   49.09   49.18   49.26   52.06   52.06   52.19   52.19   52.19
   52.19   52.04   49.24   49.33   49.33   49.33   48.96   48.77   48.53   48.27
   48.06   47.92   47.91   47.98   48.38   50.43   50.24   50.26   50.56    50.6
   50.71   51.41   52.05   52.39   51.92   53.81   54.34
   54.72   54.07   52.77   52.83   52.58   49.57   45.52   43.75   43.88   44.05
   43.72   43.79   42.86   42.88    43.6   43.61   43.61   43.61   43.62   48.09
   48.09   47.94   47.94   48.03   47.51   47.51   48.18   46.28   45.82      47
   46.89   46.95   47.08   47.55   48.37   50.42   49.78    49.6   50.55   50.22
    50.7    51.4   52.04   52.38   51.92   53.81   54.34
  4196.5  4231.5  4286.5  4301.5  4321.5  4395.8  4496.5  4601.9  4661.7  4741.7
  4795.9  4848.1  4897.2  4922.9 4944.61 4944.72 4944.83  4944.9  4945.1  4945.2
  4945.3 5048.19  5048.3 5056.99  5057.1  5057.2  5107.3  5167.9  5222.9    5275
  5312.7  5337.6  5387.7  5427.6  5497.6  5672.7  5677.7  5682.7  5697.7  5762.7
  5775.8  5800.8  5890.8  5900.8  5935.8  6105.8  6115.8
   54.72   54.07   52.78   52.84   52.59   49.58   48.37   48.26   48.19   48.68
   48.85   48.78   49.09   49.18   49.26   52.06   52.06   52.19   52.19   52.19
   52.19   52.04   49.24   49.33   49.33   49.33   48.96   48.77   48.53   48.27
   48.06   47.92   47.91   47.98   48.38   50.43   50.24   50.26   50.56    50.6
   50.71   51.41   52.05   52.39   51.92   53.81   54.34
   54.61   53.96   52.66   52.72   52.47   49.46   45.41   43.64   43.77   43.94
   43.61   43.68   42.75   42.77   43.49    43.5    43.5    43.5   43.51   47.98
   47.98   47.83   47.83   47.92    47.4    47.4   48.07   46.17   45.71   46.89
   46.78   46.84   46.97   47.44   48.26   50.31   49.67   49.49   50.44   50.11
   50.59   51.29   51.93   52.27   51.81    53.7   54.23
Pier Skew, UpSta & Num, DnSta & Num=,4962.2, 2 ,4962.2, 2 , 0 , 0 , 0 ,,
       1       1
    42.1   49.06
       1       1
   41.99   48.95
Pier Skew, UpSta & Num, DnSta & Num=,4979.0, 2 ,4979.0, 2 , 0 , 0 , 0 ,,
       1       1
   37.76   49.04
       1       1
   37.65   48.93
Pier Skew, UpSta & Num, DnSta & Num=,4995.6, 2 ,4995.6, 2 , 0 , 0 , 0 ,,
       1       1
   37.44   49.02
       1       1
   37.33   48.91
Pier Skew, UpSta & Num, DnSta & Num=,5012.5, 2 ,5012.5, 2 , 0 , 0 , 0 ,,
       1       1
   35.11   48.99
       1       1
      35   48.88
Pier Skew, UpSta & Num, DnSta & Num=,5029.5, 2 ,5029.5, 2 , 0 , 0 , 0 ,,
       1       1
   36.73   48.97
       1       1
   36.62   48.86
Abutment Skew #Up #Dn=, 2 , 2
 5040.30 5057.19
   43.66   48.03
 5040.30 5057.19
   43.55   47.92
BR Coef= 1 , 1 , 0 ,1.25, 0 ,,,0.8,0,2,0,
Wspro=,,,, 1 ,,,, 0 ,,,, 0 ,,,,-1 ,-1 ,-1 , 0 , 0 , 0 , 0 , 0
BC Design=,, 0 ,, 0 ,,,,,,
BR U #Sta/Elev= 99
  4196.5   54.72  4231.5   54.07    4241   53.85    4251   53.61    4256   53.49
    4261   53.37  4286.5   52.77  4301.5   52.83    4311   52.71    4321   52.59
  4321.5   52.58    4341   51.77  4341.5   51.75    4351   51.37    4361   50.97
    4366   50.77    4381   50.16  4395.8   49.57  4496.5   45.52  4566.5   44.38
  4601.9   43.75  4661.7   43.88  4741.7   44.05  4742.4   44.05  4795.9   43.72
    4796   43.72    4848   43.79  4848.1   43.79  4896.1   42.88  4897.2   42.86
  4922.9   42.88 4944.61    43.6 4944.72   43.61 4944.83   43.61  4944.9   43.61
 4945.01   43.62  4945.1   43.62  4945.2   43.62  4945.3   43.62  4962.2    43.3
  4965.9   41.82    4969   38.74    4979   38.77  4987.4   38.56  4995.6   38.48
  5005.2    37.7  5012.5   36.11  5019.3   36.12  5029.5   37.81  5031.1   38.95
  5032.5   41.65  5040.2   43.62  5040.3   43.66 5048.08    46.5 5048.19   46.54
  5048.3   46.58  5050.6   47.42 5056.99   47.51  5057.1   47.51  5057.2   47.51
  5107.2   48.18  5107.3   48.18  5132.4   47.39  5167.9   46.28    5168   46.28
  5221.9   45.83  5222.9   45.82  5274.4   46.99    5275      47  5296.9   46.94
  5312.7   46.89  5337.6   46.95  5387.7   47.08  5392.6   47.14  5402.6   47.25
  5427.6   47.55  5451.1   47.82  5462.6   47.96  5497.6   48.37  5513.3   48.55
  5588.3   49.43  5663.3   50.31  5668.3   50.37  5672.7   50.42  5677.7   49.78
  5682.7    49.6  5697.7   50.55  5762.7   50.22  5775.8    50.7  5800.8    51.4
  5808.3   51.45  5838.3   51.67  5890.8   52.04  5900.8   52.38  5910.9   52.25
  5935.8   51.92  5980.8   52.44  6105.8   53.81  6115.8   54.34
BR U #Mann= 6
 4196.50    0.15  4965.9   0.045  5032.5    0.15  5132.4    0.14  5296.9    0.15
  5451.1    0.14
BR U Banks=4965.90,5032.50
BR D #Sta/Elev= 99
  4196.5   54.61  4231.5   53.96    4241   53.74    4251    53.5    4256   53.38
    4261   53.26  4286.5   52.66  4301.5   52.72    4311    52.6    4321   52.48
  4321.5   52.47    4341   51.66  4341.5   51.64    4351   51.26    4361   50.86
    4366   50.66    4381   50.05  4395.8   49.46  4496.5   45.41  4566.5   44.27
  4601.9   43.64  4661.7   43.77  4741.7   43.94  4742.4   43.94  4795.9   43.61
    4796   43.61    4848   43.68  4848.1   43.68  4896.1   42.77  4897.2   42.75
  4922.9   42.77 4944.61   43.49 4944.72    43.5 4944.83    43.5  4944.9    43.5
 4945.01   43.51  4945.1   43.51  4945.2   43.51  4945.3   43.51  4962.2   43.19
  4965.9   41.71    4969   38.63    4979   38.66  4987.4   38.45  4995.6   38.37
  5005.2   37.59  5012.5      36  5019.3   36.01  5029.5    37.7  5031.1   38.84
  5032.5   41.54  5040.2   43.51  5040.3   43.55 5048.08   46.39 5048.19   46.43
  5048.3   46.47  5050.6   47.31 5056.99    47.4  5057.1    47.4  5057.2    47.4
  5107.2   48.07  5107.3   48.07  5132.4   47.28  5167.9   46.17    5168   46.17
  5221.9   45.72  5222.9   45.71  5274.4   46.88    5275   46.89  5296.9   46.83
  5312.7   46.78  5337.6   46.84  5387.7   46.97  5392.6   47.03  5402.6   47.14
  5427.6   47.44  5451.1   47.71  5462.6   47.85  5497.6   48.26  5513.3   48.44
  5588.3   49.32  5663.3    50.2  5668.3   50.26  5672.7   50.31  5677.7   49.67
  5682.7   49.49  5697.7   50.44  5762.7   50.11  5775.8   50.59  5800.8   51.29
  5808.3   51.34  5838.3   51.56  5890.8   51.93  5900.8   52.27  5910.9   52.14
  5935.8   51.81  5980.8   52.33  6105.8    53.7  6115.8   54.23
BR D #Mann= 6
 4196.50    0.15  4965.9   0.045  5032.5    0.15  5132.4    0.14  5296.9    0.15
  5451.1    0.14
BR D Banks=4965.90,5032.50

Type RM Length L Ch R = 1 ,11536.7,1466.65,1466.65,1466.65
BEGIN DESCRIPTION:
Downstream Section of Bridge/Culvert/Weir
END DESCRIPTION:
#Sta/Elev= 30
  4196.5   54.61  4321.5   52.47  4496.5   45.41  4601.9   43.64  4848.1   43.68
  4897.2   42.75  4945.3   43.51  4962.2   43.19  4965.9   41.71    4969   38.63
  4995.6   38.37  5012.5      36  5019.3   36.01  5029.5    37.7  5031.1   38.84
  5032.5   41.54  5050.6   47.31  5107.3   48.07  5132.4   47.28  5222.9   45.71
  5296.9   46.83  5451.1   47.71  5672.7   50.31  5682.7   49.49  5697.7   50.44
  5762.7   50.11  5800.8   51.29  5900.8   52.27  5935.8   51.81  6115.8   54.23
#Mann= 6 , 1 , 0
 4196.50    0.15       0  4965.9   0.045       0  5032.5    0.15       0
  5132.4    0.14       0  5296.9    0.15       0  5451.1    0.14       0
#XS Ineff= 2 , 0
       0    4935    48.7    5067       0    48.4
Bank Sta=4965.90,5032.50
Exp/Cntr=0.5,0.3

Type RM Length L Ch R = 1 ,10070.0,707,707,707
BEGIN DESCRIPTION:
Cross Section Bear Creek 14.0
END DESCRIPTION:
#Sta/Elev= 30
  3825.5   54.39  3925.5    53.7  4015.5   51.19  4205.5    50.4  4266.9   50.76
  4316.9   49.75  4356.9   47.31  4466.9   47.62  4576.9   44.66  4586.9   43.46
  4641.9   43.08  4661.9   43.77  4731.9   42.04  4826.9   41.87  4886.9   42.46
 4981.15   39.89 4988.75   37.04 5015.55   35.88 5017.95    38.4 5018.85   40.42
  5023.6   41.63  5038.6   42.23  5088.6   41.42  5208.6   42.56  5218.6   43.01
  5273.6   48.81  5288.6    51.2  5338.6   54.75  5378.6   55.37  5648.6   55.22
#Mann= 3 , 1 , 0
 3825.50    0.15       0 4981.15   0.045       0 5018.85    0.15       0
Bank Sta=4981.15,5018.85
Exp/Cntr=0.3,0.1

Type RM Length L Ch R = 1 ,9363.0,502,502,502
BEGIN DESCRIPTION:
Cross Section Bear Creek 13.0
END DESCRIPTION:
#Sta/Elev= 30
    4075   55.24    4100   54.58    4310   53.74    4390   53.73    4525   54.66
    4565   54.62  4665.9   51.66    4690   50.95    4705   49.35    4735   48.23
    4805   41.45    4920   41.07 4981.15   39.41 4988.75   36.56 5015.55    35.4
 5017.95   37.92 5018.85   39.94  5057.7   40.61  5062.7   41.49  5087.7   41.64
  5162.7   40.33  5307.7   42.66  5346.4   43.61  5402.7   44.23  5417.7   45.55
  5557.7   51.43  5577.7   52.73  5587.7   52.85  5627.7   54.86  5757.7   55.77
#Mann= 5 , 1 , 0
 4075.00     0.1       0  4665.9    0.15       0 4981.15   0.045       0
 5018.85    0.15       0  5346.4     0.1       0
Bank Sta=4981.15,5018.85
Exp/Cntr=0.3,0.1

Type RM Length L Ch R = 1 ,8861.0,722,722,722
BEGIN DESCRIPTION:
Cross Section CCX_L66
Located At: CCX_L66 CNTRL
END DESCRIPTION:
#Sta/Elev= 30
  3898.5    55.6  3968.5    54.2  4478.5   51.41  4588.5   49.08  4618.5   47.76
  4631.7   46.24  4638.5   45.46  4648.5   45.13  4703.5    44.1  4758.5      44
  4793.5   42.56  4803.5   41.51  4838.5      41  4878.5   41.18  4953.5   39.98
  4979.8   40.59  4983.5   37.09  4987.4   35.74  5014.2   34.58  5016.6    37.1
  5017.5   39.12  5036.2   40.48  5192.7   46.57  5229.2   48.41  5279.2   47.76
  5339.2   45.58  5439.2   45.61  5504.2   47.68  5639.2   54.11  5719.2   55.41
#Mann= 5 , 1 , 0
 3898.50     0.1       0  4631.7    0.15       0  4979.8   0.045       0
  5017.5    0.15       0  5192.7     0.1       0
Bank Sta=4979.80,5017.50
Exp/Cntr=0.3,0.1

Type RM Length L Ch R = 1 ,8139.0,992,992,992
BEGIN DESCRIPTION:
Cross Section Bear Creek 12.0
END DESCRIPTION:
#Sta/Elev= 30
  4217.1   55.19  4267.1      55  4342.1   54.19  4387.1   51.86  4522.1   47.34
  4532.6   47.27  4577.1   46.96  4632.1   43.58  4652.1    43.2  4722.1   43.03
  4772.1   41.97  4847.1   41.89  4917.1   42.36  4927.1   42.26  4972.1   41.08
  4977.1   40.93 4981.15   40.49 4984.85   36.99 4988.75   35.64 5015.55   34.48
 5017.95      37 5018.85   39.02  5130.4   45.34  5222.6    47.4  5310.4   49.16
  5535.4   48.34  5685.4   49.01  5770.4   52.41  5835.4   56.42  5845.4   56.57
#Mann= 6 , 1 , 0
 4217.10     0.2       0  4217.1     0.1       0  4532.6    0.15       0
 4981.15   0.045       0 5018.85    0.15       0  5222.6     0.1       0
Bank Sta=4981.15,5018.85
Exp/Cntr=0.3,0.1

Type RM Length L Ch R = 1 ,7147.0,637,637,637
BEGIN DESCRIPTION:
Cross Section Bear Creek 11.0
END DESCRIPTION:
#Sta/Elev= 30
  4386.1   54.73  4451.1   51.13  4613.9    46.2  4831.1   41.23  4931.1   41.19
 4981.15   39.37 4984.85   35.87 4988.75   34.52 5015.55   33.36 5017.95   35.88
 5018.85    35.9    5025    36.6    5080   35.95    5105   39.92    5135   40.97
  5312.3   41.15    5355    40.8    5380   43.58    5565    45.9  5650.1   49.39
  5749.5   48.36  5774.5   46.53  5794.5    42.1  5809.5      42  5869.5   47.94
  5959.5   47.06  6059.5   48.04  6419.5   47.52  6564.5   54.14  6603.9   54.65
#Mann= 7 , 1 , 0
 4386.10     0.2       0  4386.1     0.1       0  4613.9    0.15       0
 4981.15   0.045       0 5018.85    0.15       0  5312.3     0.1       0
  5650.1      10       0
Bank Sta=4981.15,5018.85
Exp/Cntr=0.3,0.1

Type RM Length L Ch R = 1 ,6510.0,623,623,623
BEGIN DESCRIPTION:
Cross Section Bear Creek 10.0
END DESCRIPTION:
#Sta/Elev= 30
  4277.1    54.1  4382.1   52.84  4547.1   46.08  4591.8    45.2  4752.1   41.22
  4782.1   39.62  4907.1   39.74 4981.15    37.2 4988.75   34.35 5015.55   33.19
 5017.95   35.71 5018.85   37.73  5030.7    39.9  5205.7   40.76  5281.8   46.74
  5355.7   46.17  5556.3   46.54  5966.3   45.71  6056.3   49.03  6100.1    49.7
  6126.3   50.08  6211.3   48.04  6241.3   48.09  6246.3   47.86  6256.3   44.08
  6261.3   43.46  6281.3    46.7  6321.3   47.09  7038.1   48.31  7174.3   53.06
#Mann= 7 , 1 , 0
 4277.10     0.2       0  4277.1     0.1       0  4591.8    0.15       0
 4981.15   0.045       0 5018.85    0.15       0  5281.8    0.15       0
  6100.1      10       0
Bank Sta=4981.15,5018.85
Exp/Cntr=0.3,0.1

Type RM Length L Ch R = 1 ,5887.0,640,640,640
BEGIN DESCRIPTION:
Cross Section Bear Creek 9.0
END DESCRIPTION:
#Sta/Elev= 30
  3970.2   52.03  4000.2   50.63  4120.2   47.84  4140.2   47.92  4195.2   45.77
  4255.2   46.94  4339.4   45.56  4495.2   40.53  4585.2   39.36  4833.7   39.01
  4888.7   37.58 4981.15   37.56 4988.75   34.18 5015.55   33.02 5017.95   35.54
 5018.85   37.56  5113.7   40.07  5173.7   47.37  5363.7   46.83  5400.2   46.66
  5865.6   47.09  6270.6   44.51  6315.6   44.83  6475.6   48.26  6665.6   47.29
  6720.6   46.07  6920.6   47.37  7350.6   46.99  7440.6   52.52  7520.6   56.23
#Mann= 7 , 1 , 0
 3970.20     0.2       0  3970.2     0.1       0  4339.4    0.15       0
 4981.15   0.045       0 5018.85    0.15       0  5363.7     0.1       0
  5400.2      10       0
Bank Sta=4981.15,5018.85
Exp/Cntr=0.3,0.1

Type RM Length L Ch R = 1 ,5247.0,386,386,386
BEGIN DESCRIPTION:
Cross Section Bear Creek 8.0
END DESCRIPTION:
#Sta/Elev= 30
  3537.9   50.74  3577.9   49.61  3922.9    48.7  4272.9    45.6  4499.9   49.03
  4562.9   48.03    4666   41.49  4721.3   38.34  4901.3   35.62 4981.15   36.28
 4988.75   33.93 5015.55   32.77 5018.85   37.31  5100.4   39.46  5150.4   44.49
  5165.4   44.51  5175.4   46.78  5225.4   49.21  5249.9   48.76  5325.4   47.82
  5340.4   46.21  5855.4   45.74  5945.4   47.08  6520.4    45.5  6700.4   46.71
  6740.4    48.2  6915.4   45.89  7345.4   45.91  7480.4   52.43    7554   53.77
#Mann= 7 , 1 , 0
 3537.90     0.2       0  3537.9      10       0  4499.9     0.1       0
    4666    0.15       0 4981.15   0.045       0 5018.85    0.15       0
  5249.9      10       0
Bank Sta=4981.15,5018.85
Exp/Cntr=0.3,0.1

Type RM Length L Ch R = 1 ,4861.0,1114,1114,1114
BEGIN DESCRIPTION:
Cross Section Bear Creek 7.0
END DESCRIPTION:
#Sta/Elev= 30
    3499    50.9    3584   49.67    3629   45.36    3659   43.76    3829   42.18
    3904   42.26    3984   46.54    4104   48.01    4289   46.14    4349    46.3
    4425   49.89    4539   47.45  4590.4   44.11    4619    42.9  4709.4   43.44
  4804.4   38.86  4849.4   39.31  4894.4   37.03 4981.15   36.77 4988.75   33.92
 5015.55   32.76 5017.95   35.28 5018.85    37.3  5074.4   40.49  5134.4   45.67
  5484.4   43.46  5581.6   43.53  5994.3   45.85  7339.3   49.68  7463.2   52.59
#Mann= 7 , 1 , 0
 3499.00      10       0    4425     0.1       0  4590.4    0.15       0
 4981.15   0.045       0 5018.85    0.15       0  5581.6     0.1       0
  7463.2     0.2       0
Bank Sta=4981.15,5018.85
Exp/Cntr=0.3,0.1

Type RM Length L Ch R = 1 ,3747.0,379,379,379
BEGIN DESCRIPTION:
Cross Section Bear Creek 6.0
END DESCRIPTION:
#Sta/Elev= 30
  3378.8   51.83  3478.8   48.25  3523.8   43.53  3583.8   40.35  3748.8   47.54
  3849.8   48.38    3902   47.85    3957   44.11    4142   45.81    4192   41.46
  4268.4   39.64    4417   41.06    4477   38.25    4617   42.48    4692   39.46
    4892   39.89 4981.15   36.75 4988.75    33.9 5015.55   32.74 5018.85   37.28
  5050.5   38.04  5100.5   42.49  5245.5   42.62  5385.5    45.9  5565.2   44.76
  5670.5   43.58  6149.8   47.28  6765.5   46.63  6815.5   50.38  6901.5   52.92
#Mann= 7 , 1 , 0
 3378.80      10       0  3849.8     0.1       0  4268.4    0.15       0
 4981.15   0.045       0 5018.85    0.15       0  5565.2     0.1       0
  6149.8      10       0
Bank Sta=4981.15,5018.85
Exp/Cntr=0.3,0.1

Type RM Length L Ch R = 1 ,3368.0,394,394,394
BEGIN DESCRIPTION:
Cross Section Bear Creek 5.0
END DESCRIPTION:
#Sta/Elev= 30
    3284   49.92    3314   48.78    3409   40.44    3459   41.03    3469    42.1
  3984.7   46.72    4269   43.91    4524   42.35  4681.5    42.2    4849   41.99
    4929   40.31    4934   39.44 4981.15   36.74 4988.75   33.89 5015.55   32.73
 5017.95   35.25 5018.85   37.27    5080   41.07    5150   42.55    5210   45.15
    5245   45.48    5265   46.87  5299.7   47.28    5315   47.46    5380   44.43
    5495   42.61    5720   45.14    5880   48.51    6730      51  6745.2   52.73
#Mann= 6 , 1 , 0
 3284.00      10       0  3984.7     0.1       0  4681.5    0.15       0
 4981.15   0.045       0 5018.85    0.15       0  5299.7      10       0
Bank Sta=4981.15,5018.85
Exp/Cntr=0.3,0.1

Type RM Length L Ch R = 1 ,2974.0,769,769,769
BEGIN DESCRIPTION:
Cross Section Bear Creek 4.0
END DESCRIPTION:
#Sta/Elev= 30
    3072   51.28    3192   42.68    3367   42.95    3477   45.45    3747   47.01
  3819.9   46.77    4387   43.89  4459.8   38.72    4597   38.35    4642   39.92
    4717   41.07    4817   42.28    4892    42.3  4959.8   41.33  4979.8   40.46
 4981.15   38.76 4984.85   35.26 4988.75   33.91 5015.55   32.75 5017.95   35.27
 5018.85   37.29  5059.8   43.69  5069.8   44.68  5104.8   46.53  5237.5   46.85
  5307.8   47.21  5317.8   47.81  5417.8   47.77  5502.8   48.87  5562.8   51.18
#Mann= 6 , 1 , 0
 3072.00      10       0  3819.9     0.1       0  4459.8    0.15       0
 4981.15   0.045       0 5018.85    0.15       0  5237.5     0.1       0
Bank Sta=4981.15,5018.85
Exp/Cntr=0.3,0.1

Type RM Length L Ch R = 1 ,2205.0,573,573,573
BEGIN DESCRIPTION:
Cross Section Bear Creek 3.0
END DESCRIPTION:
#Sta/Elev= 30
    3785   52.91    3845   48.91    3995   47.04    4100   47.11    4355   45.32
  4599.8   46.99  4837.1   43.86    4920   44.03 4981.15   38.32 4984.85   34.82
 4988.75   33.47 5015.55   32.31 5017.95   34.83 5018.85   36.85  5116.5   39.77
  5121.5   41.65  5206.5   44.41  5231.5   43.37  5301.5   43.14  5356.5    39.4
  5451.5   39.57    5474   40.54  5521.5   42.37  5531.5   43.77  5551.5    42.3
  5586.5   42.32  5806.5   47.71  5871.5   46.34  5929.7   47.81  6036.9   51.11
#Mann= 7 , 1 , 0
 3785.00      10       0  4599.8     0.1       0  4837.1    0.15       0
 4981.15   0.045       0 5018.85    0.15       0    5474     0.1       0
  5929.7     0.2       0
Bank Sta=4981.15,5018.85
Exp/Cntr=0.3,0.1

Type RM Length L Ch R = 1 ,1632.0,0,0,0
BEGIN DESCRIPTION:
Cross Section Bear Creek 2.0
END DESCRIPTION:
#Sta/Elev= 30
  3612.4    50.9  4197.4   47.75  4352.4    47.2  4512.4   47.56  4562.4      46
  4577.4   44.86    4587   44.76  4722.4   43.39  4787.4   41.23  4872.4   41.17
  4887.4      41  4942.4   39.66 4981.15   37.99 4984.85   34.49 4988.75   33.14
 5015.55   31.98 5017.95    34.5 5018.85   36.52  5022.4   36.76  5043.5   37.12
  5073.5   39.61  5138.5   41.18  5265.4   43.48  5333.5   44.72  5363.5   46.44
  5383.5   46.37  5708.5   46.95  5778.5   50.29  5793.5   51.37    5835   52.14
#Mann= 6 , 1 , 0
 3612.40     0.1       0    4587    0.15       0 4981.15   0.045       0
 5018.85    0.15       0  5265.4     0.1       0    5835     0.2       0
Bank Sta=4981.15,5018.85
Exp/Cntr=0.3,0.1

Chan Stop Cuts=-1
