--- DTL_Cow_Branch.prj (project) ---

Proj Title=DTL_Cow_Branch
Current Plan=p01
Default Exp/Contr=0.3,0.1
English Units
Geom File=g01
Flow File=f01
Flow File=f02
Plan File=p01
Plan File=p02
Y Axis Title=Elevation
X Axis Title(PF)=Main Channel Distance
X Axis Title(XS)=Station
BEGIN DESCRIPTION:
END DESCRIPTION:
DSS Export Rating Curves= 0
DSS Export Rating Curve Sorted= 0
DSS Export Volume Flow Curves= 0
DXF OffsetX= 0
DXF OffsetY= 0
DXF ScaleX= 1
DXF ScaleY= 10

--- DTL_Cow_Branch.p01 (plan) ---

Plan Title=DTL_Cow_Branch
Program Version=4.00
Short Identifier=Multi Profile
Geom File=g01
Flow File=f01
Subcritical Flow
K Sum by GR= 0
Std Step Tol= 0.01
Critical Tol= 0.01
Num of Std Step Trials= 20
Max Error Tol= 0.3
Flow Tol Ratio= 0.001
Split Flow NTrial= 30
Split Flow Tol= 0.02
Split Flow Ratio= 0.02
Log Output Level= 0
Friction Slope Method= 1
Unsteady Friction Slope Method= 2
Unsteady Bridges Friction Slope Method= 1
Parabolic Critical Depth
Global Vel Dist= 0 , 0 , 0
Global Log Level= 0
CheckData=True
Encroach Param=-1 ,10,10, 2
Encroach River=Cow Branch
Encroach Reach=Main
Encroach Node=21222
       1     255     290
Encroach Node=21002
       1     299  349.96
Encroach Node=20423
       1     355     412
Encroach Node=20072
       1     440     515
Encroach Node=19891
       1     585     661
Encroach Node=19774
       1     595     669
Encroach Node=19576
       1     415     445
Encroach Node=18989
       1     320     375
Encroach Node=18593
       1     270     335
Encroach Node=18036
       1     395     460
Encroach Node=17554
       1     380     555
Encroach Node=17222
       1     385     530
Encroach Node=16772
       1     435     515
Encroach Node=15835
       1     385     475
Encroach Node=15381
       1     550     640
Encroach Node=15130
       1     400     480
Encroach Node=14647
       1     390     470
Encroach Node=14187
       1     340     415
Encroach Node=13839
       1     490     560
Encroach Node=13571
       1     500     575
Encroach Node=13170
       1     320     420
Encroach Node=12622
       1     600     700
Encroach Node=11707
       1     445     550
Encroach Node=11070
       1     320     420
Encroach Node=10425
       1     290     385
Encroach Node=10016
       1     495     575
Encroach Node=9822
       1  667.38  710.63
Encroach Node=9742
       1  671.57 700.805
Encroach Node=9537
       1     380     440
Encroach Node=9012
       1     590     663
Encroach Node=8630
       1     330     420
Encroach Node=8141
       1     440     530
Encroach Node=7924
       1     400     490
Encroach Node=7292
       1     500     595
Encroach Node=6747
       1     493   593.1
Encroach Node=6417
       1     605     705
Encroach Node=6032
       1     490     570
Encroach Node=5364
       1     500     580
Encroach Node=4871
       1     360     470
Encroach Node=4234
       1     545     675
Encroach Node=3479
       1  292.16     415
Encroach Node=2845
       1     360     425
Encroach Node=2690
       1  818.04  861.96
Encroach Node=2559
       1  842.76  881.96
Encroach Node=2396
       1  617.57  650.27
Encroach Node=2307
       1     580  618.53
Encroach Node=1765
       1     280     335
Encroach Node=1379
       1     490     550
Computation Interval=1HOUR
Output Interval=1HOUR
Run HTab= 0
Run UNet= 0
Run PostProcess= 0
Run WQNet= 0
UNET Theta= 1
UNET Theta Warmup= 1
UNET ZTol= 0.02
UNET ZSATol= 0.05
UNET MxIter= 20
UNET MaxInSteps= 0
UNET DtIC= 0
UNET DtMin= 0
UNET MaxCRTS= 20
UNET WFStab= 2
UNET SFStab= 1
UNET WFX= 1
UNET SFX= 1
UNET DSS MLevel= 4
UNET DZMax Abort= 100
UNET Convert EG Bridges= 0
UNET Use Existing IB Tables=-1
UNET Froude Reduction=False
UNET Froude Limit= 1
UNET Froude Power= 10
UNET Time Slicing=0,0, 5
Instantaneous Interval=1HOUR
Write IC File= 0
Echo Input=False
Echo Output=False
Write Detailed= 0
Detailed Automatic Start=False, 10
WQ ULTIMATE=-1
WQ Max Comp Step=1HOUR
WQ Output Interval=15MIN
WQ Output Selected Increments= 0
WQ Output face flow=0
WQ Output face velocity=0
WQ Output face area=0
WQ Output face dispersion=0
WQ Output cell volume=0
WQ Output cell surface area=0
WQ Output cell continuity=0
WQ Output face conc=0
WQ Output face dconc_dx=0
WQ Output face courant=0
WQ Output face peclet=0
WQ Output face adv mass=0
WQ Output face disp mass=0
WQ Output cell mass=0
WQ Output cell source sink temp=0
WQ Output cell source sink nsm=0
WQ Output MaxMinRange=-1
WQ Daily Max Min Mean=-1
WQ Daily Range=0
WQ Daily Time=0
WQ Create Restart=0
WQ Fixed Restart=0
WQ System Summary=False
Sorting and Armoring Iterations= 10
XS Update Threshold= 0.02
Hydraulics Update Threshold= 0.02
Energy Slope Method= 1
Volume Change Method= 0
XS Weighting Method= 0
Number of US Weighted Cross Sections= 1
Number of DS Weighted Cross Sections= 1
Upstream XS Weight=0.25
Main XS Weight=0.5
Downstream XS Weight=0.25
Number of DS XS's Weighted with US Boundary= 1
Upstream Boundary Weight= 1
Weight of XSs Associated with US Boundary= 0
Number of US XS's Weighted with DS Boundary= 1
Downstream Boundary Weight= 0.5
Weight of XSs Associated with DS Boundary= 0.5
Sediment Output Level= 4
Mass or Volume Output= 0
Output Increment Type= 1
Profile and TS Output Increment= 10
XS Output Flag= 0
XS Output Increment= 10
Disregard all LS=0
Disregard all Conn=0
Disregard all Breaches=0
Disregard all Pumps=0

--- DTL_Cow_Branch.p02 (plan) ---

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Plan Title=DTL_Cow_Branch_Future
Short Identifier=Future
Geom File=g01
Flow File=f02
Encroach Param=-1 ,0,0, 0

--- DTL_Cow_Branch.f01 (steady flow) ---

Flow Title=DTL_Cow_Branch
Program Version=4.00
Number of Profiles= 6
Profile Names=100-yr,FW,10-yr,25-yr,50-yr,500-yr
River Rch & RM=Cow Branch,Main            ,21222
     470     470     190     280     370     770
River Rch & RM=Cow Branch,Main            ,16772
     670     670     280     410     530    1090
River Rch & RM=Cow Branch,Main            ,12622
     850     850     360     530     680    1370
River Rch & RM=Cow Branch,Main            ,9012
    1000    1000     430     620     800    1590
River Rch & RM=Cow Branch,Main            ,4871
    1070    1070     460     670     850    1690
Boundary for River Rch & Prof#=Cow Branch,Main            , 1
Up Type= 0
Dn Type= 3
Dn Slope=0.00203
Boundary for River Rch & Prof#=Cow Branch,Main            , 2
Up Type= 0
Dn Type= 3
Dn Slope=0.00203
Boundary for River Rch & Prof#=Cow Branch,Main            , 3
Up Type= 0
Dn Type= 3
Dn Slope=0.00203
Boundary for River Rch & Prof#=Cow Branch,Main            , 4
Up Type= 0
Dn Type= 3
Dn Slope=0.00203
Boundary for River Rch & Prof#=Cow Branch,Main            , 5
Up Type= 0
Dn Type= 3
Dn Slope=0.00203
Boundary for River Rch & Prof#=Cow Branch,Main            , 6
Up Type= 0
Dn Type= 3
Dn Slope=0.00203
DSS Import GetInterval= 0
DSS Import GetPeak= 0
DSS Import FillOption= 0

--- DTL_Cow_Branch.f02 (steady flow) ---

Flow Title=DTL_Cow_Branch_Future
Program Version=4.00
Number of Profiles= 3
Profile Names=100-yr 10%,100-yr 20%,100-yr 35%
River Rch & RM=Cow Branch,Main            ,21222
     830    1060    1300
River Rch & RM=Cow Branch,Main            ,16772
    1180    1510    1850
River Rch & RM=Cow Branch,Main            ,12622
    1480    1900    2320
River Rch & RM=Cow Branch,Main            ,9012
    1730    2210    2700
River Rch & RM=Cow Branch,Main            ,4871
    1830    2350    2870
Boundary for River Rch & Prof#=Cow Branch,Main            , 1
Up Type= 0
Dn Type= 3
Dn Slope=0.00203
Boundary for River Rch & Prof#=Cow Branch,Main            , 2
Up Type= 0
Dn Type= 3
Dn Slope=0.00203
Boundary for River Rch & Prof#=Cow Branch,Main            , 3
Up Type= 0
Dn Type= 3
Dn Slope=0.00203
DSS Import GetInterval= 0
DSS Import GetPeak= 0
DSS Import FillOption= 0

--- DTL_Cow_Branch.g01 (geometry) ---

Geom Title=DTL_Cow_Branch
Program Version=4.00

River Reach=Cow Branch      ,Main
Reach XY= 30
2357196.36505805618793.3534543072357170.84945469619023.683495983
2356846.04271923619439.5188706222356997.04839176619965.940333858
2357200.50272346620365.6663136782357801.15382023620657.371725738
2358134.23588648621216.6461682622358131.47744285621619.378935754
2357796.32654391622091.0727935582357620.29726121623946.542990446
2358070.10207245624737.1098292472358017.00203291625663.257272303
2358354.22176458626365.2811717692358634.89340223629063.728636101
2358905.91048718629415.4301967622359082.45087838630355.369857848
2359270.71465501630607.7674484252359256.23282604631389.786212713
2359406.56800291631651.8383559292359278.98998582632496.611712411
2359387.25889762632613.1559550322359219.68344815632802.109342515
2359372.08745775633451.0332024692359089.34698743634043.408968329
2359242.44060794634280.6351190362359381.05239949635208.851394773
2359246.57827334635401.9424476772359312.09130916635686.751750723
2359171.41068494636459.8055732552359351.34257299637095.575231478

Type RM Length L Ch R = 1 ,21222   ,192.17,219.12,284.4
XS GIS Cut Line= 3
2356923.15454826618798.2531949432357196.36505805618793.353454307
 2357618.6284703618767.845009103
#Sta/Elev= 30
       0  121.26   95.05  120.89  112.63  121.16  154.02120.8876  180.56  120.68
  197.34  120.91  217.51  119.78  234.62   117.5  261.81  113.03  263.41  112.89
   265.2  111.99  271.85   110.4  280.17  111.99  283.32  113.07  289.42  114.06
  318.27  112.34  332.06  112.05  361.92  111.58  388.15  112.23  411.74   113.7
  447.73  113.89     492   116.2   541.9   117.7  565.82   118.7  593.07  120.27
  604.36  122.58  622.45  122.53  630.87   122.8  649.77  122.62  696.29  123.19
#Mann= 5 ,-1 , 0
       0    .045       0  154.02    .085       0  261.81     .05       0
  283.32    .075       0  332.06    .045       0
#XS Ineff= 2 , 0
       0                     290       0  116.13
Permanent Ineff=
       F       F
Bank Sta=261.81,283.32
XS Rating Curve= 0 ,0
Exp/Cntr=0.3,0.1

Type RM Length L Ch R = 1 ,21002   ,659.57,579.7,479.83
XS GIS Cut Line= 2
2356918.62293041618839.0377558082357539.61971966619243.651664098
#Sta/Elev= 30
       0  121.18   19.14  121.32   50.29  121.02   83.86  121.21  120.22  120.89
   141.2  121.27  175.24  121.71  240.13  116.53  285.22  111.86  289.29  112.33
  301.04  110.39  302.49  110.04  321.44  108.82  339.09  110.13  347.82  110.42
  379.86  110.97  388.67  111.33  420.64  113.63  426.64  113.84  439.18   113.6
  460.43  113.88  480.45  114.22  501.49  115.01     523  115.41  583.39  117.76
  591.48  118.36  603.94  118.59  647.98  120.45  690.23  121.86  741.18  122.91
#Mann= 5 ,-1 , 0
       0    .045       0   141.2    .085       0  301.04     .05       0
  347.82    .075       0  379.86    .045       0
Bank Sta=301.04,347.82
XS Rating Curve= 0 ,0
Exp/Cntr=0.3,0.1

Type RM Length L Ch R = 1 ,20423   ,360.53,351.06,308.98
XS GIS Cut Line= 3
2356469.42230764619496.8680160342357028.40934874 619456.25784637
2357286.40336767 619513.58985059
#Sta/Elev= 30
       0   122.5   68.73  121.32   95.37   120.5  126.19  116.81   186.3  114.67
  237.03   113.4  257.16  112.51   287.6   111.2  334.35  109.65  344.69  109.64
  366.08  107.39  377.18  105.75  380.71  105.51  391.67  107.38  393.78  107.59
  407.59  107.16   411.7  107.69  444.39  107.93  470.21  107.67  502.97  108.93
  535.12  111.83  578.87  114.31  613.08  117.03  688.45  122.12  712.75  122.47
  740.57  122.19  758.09  122.25  789.45  122.61  804.29  122.52  824.75  123.06
#Mann= 5 ,-1 , 0
       0     .04       0  257.16    .085       0  366.08     .05       0
  391.67    .085       0  712.75     .04       0
Bank Sta=366.08,391.67
XS Rating Curve= 0 ,0
Exp/Cntr=0.3,0.1

Type RM Length L Ch R = 1 ,20072   ,202.53,180.51,180.16
XS GIS Cut Line= 2
2356490.92180921619924.4692141412357291.18103468619697.530030772
#Sta/Elev= 30
       0  124.46   36.04  123.92  106.81  121.77  144.73  120.99  180.48  115.54
  189.83  115.59  215.52  114.79  268.92  112.34  298.33  110.41  317.67  109.58
  333.82  108.99  366.32  108.54  371.91  108.08  379.92  108.55  388.57  106.87
  420.77  105.35  436.59  105.66  463.94  104.96  481.48  105.21  491.89   103.6
  498.21  103.97  502.59  105.22  544.79   107.4  592.38  111.74  607.53  112.51
   698.4  118.56  751.52  122.65  763.94  123.23  776.58  123.78  831.81  123.74
#Mann= 5 ,-1 , 0
       0     .04       0  317.67    .085       0  481.48     .05       0
  502.59    .085       0  763.94     .04       0
Bank Sta=481.48,502.59
XS Rating Curve= 0 ,0
Exp/Cntr=0.5,0.3

Type RM Length L Ch R = 1 ,19891   ,118.39,117.2,113.24
BEGIN DESCRIPTION:
Surveyed Section
END DESCRIPTION:
XS GIS Cut Line= 6
2356372.47931616620107.1970738922356741.34705006 620072.83266075
2356848.91905379620041.6933965092357030.57960002619934.617100015
2357226.83648804619932.7059716582357294.77670096619910.059234023
#Sta/Elev= 30
       0  124.86  114.94  123.84   196.9  122.29  277.54  120.14  307.86  119.82
  329.77  117.26  361.21  115.65  388.94  113.27  418.85  111.83  450.86  109.52
   469.6  109.04     528  108.02 564.345  105.43  614.32  105.25 647.165  104.13
  647.65  103.42  649.16  102.57  651.72  102.61 652.319  104.11  727.67  109.15
  747.02  108.78  788.64   110.5  797.44  110.36  811.73  111.18  827.43  111.42
  852.48  112.64  892.85  115.87  907.84  118.09  935.24   120.1  964.47  120.84
#Mann= 5 ,-1 , 0
       0     .04       0   469.6    .085       0 647.165     .05       0
 652.319    .085       0  935.24     .04       0
#XS Ineff= 2 , 0
       0     637  107.65     661       0   109.5
Permanent Ineff=
       F       F
Bank Sta=647.165,652.319
XS Rating Curve= 0 ,0
Exp/Cntr=0.5,0.3

Type RM Length L Ch R = 2 ,19833   ,,,
BEGIN DESCRIPTION:
Shine Road (+/- 0.25 mi)
END DESCRIPTION:
Bridge Culvert--1,0,-1,-1, 0
Deck Dist Width WeirC Skew NumUp NumDn MinLoCord MaxHiCord MaxSubmerge Is_Ogee
51.5,9.5,2.6,0, 41, 41, , , 0.98, 0, 1,1,,
       0    20.5   70.48    92.8  149.74  171.38  202.98  248.86  278.33  298.11
  315.76   339.1  345.92  377.64  408.46  419.96   421.3  427.15  438.06  453.72
   480.3  493.23  512.96 551.643 586.353 623.208 655.754 697.254 735.415  751.47
  775.64  810.39  830.06  830.63  850.82  880.75   925.5  940.02   945.7  958.93
  969.06
  124.93  125.04  124.26   123.5  122.08  121.82     121  120.08  119.63  118.78
  116.88  113.85  113.64  112.42  110.32  109.78  109.75  109.59  109.33  109.07
  108.85  108.67  108.09  107.65  107.84  108.49  109.22  109.64  110.15  110.27
  110.26  113.52  113.52  113.61   115.3  117.42  119.15  119.27  119.27   119.1
   119.1
                                                                                
                                                                                
                                                                                
                                                                                
        
       0    20.5   70.48    92.8  149.74  171.38  202.98  248.86  278.33  298.11
  315.76   339.1  345.92  377.64  408.46  419.96   421.3  427.15  438.06  453.72
   480.3  493.23  512.96 551.643 586.353 623.208 655.754 697.254 735.415  751.47
  775.64  810.39  830.06  830.63  850.82  880.75   925.5  940.02   945.7  958.93
  969.06
  124.93  125.04  124.26   123.5  122.08  121.82     121  120.08  119.63  118.78
  116.88  113.85  113.64  112.42  110.32  109.78  109.75  109.59  109.33  109.07
  108.85  108.67  108.09  107.65  107.84  108.49  109.22  109.64  110.15  110.27
  110.26  113.52  113.52  113.61   115.3  117.42  119.15  119.27  119.27   119.1
   119.1
                                                                                
                                                                                
                                                                                
                                                                                
        
BR Coef= 1 , 1 , 0 ,1.25, 0 ,,,0.8,0,2,0,
WSPro=,,,, 1 ,,,, 0 ,,,, 0 ,,,,-1 ,-1 ,-1 , 0 , 0 , 0 , 0 , 0
Culvert=1,4,,21,0.024,0.5,1,2,1,102.19,649,102,657,Culvert #1  , 0 ,46.5
Culvert Bottom n=0.024
BC Design=,, 0 ,, 0 ,,,,,,
BC Use User HTab Curves=0
BC User HTab FreeFlow(D)= 0

Type RM Length L Ch R = 1 ,19774   ,177.31,198.18,159.52
BEGIN DESCRIPTION:
Surveyed Section
END DESCRIPTION:
XS GIS Cut Line= 6
2356422.34105623620216.2696302092356763.99378772620183.235506698
2357006.96910001620098.007499993    2357089.8928620035.837700009
2357245.23696235620038.8625543122357345.82203303619999.163303822
#Sta/Elev= 30
       0  121.83   24.81  121.86   53.41  121.29  173.97  116.11  197.22  115.39
  257.43  114.54  326.26  111.71  447.03109.4455  517.29  108.09  537.65  106.12
  582.43  106.26  597.02  106.07 601.262  105.52  652.48  105.13 654.257  103.78
  655.55  102.06  658.62  102.03 659.768  103.95 664.015  105.24 705.303  106.61
  713.25  107.49  749.99  109.71  773.13  109.92  782.09  110.44  788.11   111.4
  822.87  112.97  868.49  116.11  895.89  117.11  941.54  118.08  969.06  117.76
#Mann= 5 ,-1 , 0
       0     .04       0  447.03    .085       0 654.257     .05       0
 659.768    .085       0  895.89     .04       0
#XS Ineff= 3 ,-1
       0     250     120                             669    1000  109.22
Permanent Ineff=
       F       F       F
Bank Sta=654.257,659.768
XS Rating Curve= 0 ,0
Exp/Cntr=0.5,0.3

Type RM Length L Ch R = 1 ,19576   ,640.72,586.72,499.22
XS GIS Cut Line= 4
2356714.70012614620404.7117306292357054.86282416620270.814687401
2357222.94408005620189.4279740452357421.63251424620019.524211496
#Sta/Elev= 30
       0  119.37   91.29  118.98  114.18  118.49  172.44  116.14  206.85  114.46
  258.96  111.05  277.97  110.56  305.95   109.5  331.12   107.9  352.83  107.57
  378.76  105.19  402.31  103.56  420.21  103.22   432.5  101.73  441.49   103.2
  454.76  104.02  492.77  103.19  530.26  103.58  547.86  105.25   584.3  110.02
  595.36  110.22  612.94  111.68  635.88  114.38  647.92  114.44  665.84  115.46
   683.7  115.93  699.17  115.27  748.12  116.12  771.23  116.12  813.74  116.73
#Mann= 5 ,-1 , 0
       0     .04       0  277.97    .085       0  420.21     .05       0
  441.49    .085       0  699.17     .04       0
Bank Sta=420.21,441.49
XS Rating Curve= 0 ,0
Exp/Cntr=0.3,0.1

Type RM Length L Ch R = 1 ,18989   ,327.46,396.49,414.11
XS GIS Cut Line= 2
2357374.05052654620882.7974161652357768.30128142620196.257308528
#Sta/Elev= 30
       0  118.52   10.43  117.74   31.72   116.8   55.58  115.11   74.47  115.41
   82.34  114.37   95.99   113.4  127.43  113.35   132.6  113.09  190.93   109.8
  234.15  105.41  259.12  104.14  278.43  103.07  307.05  100.92   333.4   99.85
  343.94   97.79  353.44   99.33  359.32   99.84  379.35   100.6  442.12  100.48
   486.1  104.23  525.55  107.23  542.03  108.95  573.81  111.53  617.06  112.32
  642.43  113.79  667.08  112.91  683.51  112.81  731.82  114.85  791.69  115.85
#Mann= 7 ,-1 , 0
       0    .085       0   55.58     .09       0  259.12    .085       0
   333.4     .05       0  359.32    .085       0   486.1    .075       0
  667.08     .04       0
Bank Sta=333.4,359.32
XS Rating Curve= 0 ,0
Exp/Cntr=0.3,0.1

Type RM Length L Ch R = 1 ,18593   ,503.87,557.1,581.5
XS GIS Cut Line= 3
2357616.49208273620980.2272004042358096.96661048620565.620363787
2358128.56490226620497.609897017
#Sta/Elev= 30
       0  116.84   23.61  116.15   77.26  112.62   87.69  112.27  110.92  109.88
  124.43  107.84     163  103.05  208.61   98.94  237.62   97.95     264   98.15
  313.02   97.36  320.76   95.79  326.95   97.04  332.65    97.4  357.22    98.7
  386.53  101.24  412.43  102.55  429.66  103.44  447.63  105.25  460.23  107.22
  471.41  107.69  492.58  109.66  513.34  110.96  530.45  111.13  547.43  111.95
  570.61  112.58  609.28  113.06  631.66  113.98  651.36  113.96  709.62  115.28
#Mann= 5 ,-1 , 0
       0     .09       0     163    .085       0  313.02     .05       0
  332.65     .09       0  412.43    .075       0
Bank Sta=313.02,332.65
XS Rating Curve= 0 ,0
Exp/Cntr=0.3,0.1

Type RM Length L Ch R = 1 ,18036   ,428.91,481.31,555.96
XS GIS Cut Line= 4
2357720.71929379 621209.073902952358017.34917347621253.426555529
2358563.61325505621111.8844453392358690.48551844621127.504781261
#Sta/Elev= 30
       0  113.79   61.86  112.49   95.44   110.8  130.53  111.01  174.75  109.64
  227.16  109.31  284.66  108.04  309.15  106.71  321.68  106.62  331.17  105.77
  363.78  101.47   377.3   97.28  401.59   95.86   419.1   95.96  428.23   95.62
  431.15   95.95   499.7   96.94  526.08   96.78   541.2   97.73   578.7   97.25
  608.69   99.71  627.77  100.32  687.98  104.72  710.91  105.99  717.01  105.63
  745.68   106.2  793.74  108.77  814.28  109.43  876.48  111.26  992.06  113.75
#Mann= 4 ,-1 , 0
       0     .09       0   419.1     .05       0  431.15     .09       0
  710.91     .04       0
#XS Ineff= 2 , 0
                          542.89           98.84
Permanent Ineff=
       F       F
Bank Sta=419.1,431.15
XS Rating Curve= 0 ,0
Exp/Cntr=0.3,0.1

Type RM Length L Ch R = 1 ,17554   ,327.39,332.4,326.96
XS GIS Cut Line= 5
2357656.33241129621524.0474019942358032.42764585 621657.39025788
2358206.79907276621751.4140665232358263.21335797 621831.76168482
2358548.70383145622173.666443512
#Sta/Elev= 30
       0  108.45    34.5  108.17   50.65  108.47  122.92  107.64   168.9  106.53
  206.91  105.91  234.78  105.95  261.23  105.34   335.8   99.63  376.67   96.01
  382.65   96.06  397.05   95.46  404.99    95.6  409.15   96.11  432.07   96.36
  465.45   95.96  553.49    96.4  569.02   96.87  589.06   98.65  621.38  103.02
  631.29  103.24  641.51   102.8  664.59  103.15  695.31  103.35  724.04  104.07
  832.64  104.92  890.58  105.93  901.13  106.46 1007.65  108.85 1140.74  113.16
#Mann= 6 ,-1 , 0
       0     .04       0  261.23     .09       0  382.65    .032       0
  553.49    .032       0  553.49    .085       0  664.59     .04       0
Bank Sta=382.65,553.49
XS Rating Curve= 0 ,0
Exp/Cntr=0.3,0.1

Type RM Length L Ch R = 1 ,17222   ,463.99,449.68,376.16
XS GIS Cut Line= 4
2357580.23913975621650.9066455072357764.03241029621877.918827251
2358076.87526447622052.2902541612358497.41811764622233.499776289
#Sta/Elev= 30
       0  109.03   69.58  109.41  101.32  108.49  107.27   108.8  174.06  108.59
  211.77  107.92  291.76  103.15  313.26   100.3  321.08   98.58  351.85   93.54
  396.57   92.66  417.39   93.04  430.97    92.5  444.17   90.84   451.6   92.39
  456.51   92.51  469.66   92.52  479.05   93.22  493.54   92.57     527   94.09
  557.22   94.81  576.76   96.12  591.65   96.03  599.79   97.12   623.2   98.73
  645.17   99.23  688.92  100.34  790.86  104.22  940.78  107.78 1108.17   113.1
#Mann= 5 ,-1 , 0
       0     .09       0  211.77     .07       0  430.97     .05       0
  456.51    .085       0  645.17     .04       0
Bank Sta=430.97,456.51
XS Rating Curve= 0 ,0
Exp/Cntr=0.3,0.1

Type RM Length L Ch R = 1 ,16772   ,888.26,937.15,954.21
XS GIS Cut Line= 4
2357312.87368526622321.5860905652357400.31403689 622348.16631408
2358015.13757804622361.4358869052358214.66564184622439.408155248
#Sta/Elev= 30
       0  116.54  124.61  113.28  146.33  111.74   185.7  110.31  222.93  105.91
  234.29  105.09  243.39  103.47  310.44   97.06  339.08   95.33   363.5   92.91
  380.66    93.3  389.74    93.6  456.55   92.92  463.84   91.75  471.01   89.32
  479.35   91.72  493.38   92.84     523    93.2  536.41   92.67  554.54   93.36
  573.99   92.55  595.25   95.32  611.51   98.12  618.35    98.5  667.01  104.98
  677.06  104.89  696.79  105.81   739.6  108.26  756.03  108.67  920.58  111.28
#Mann= 6 ,-1 , 0
       0     .09       0  380.66     .07       0  463.84     .05       0
  479.35    .085       0  595.25    .075       0  696.79     .04       0
Bank Sta=463.84,479.35
XS Rating Curve= 0 ,0
Exp/Cntr=0.3,0.1

Type RM Length L Ch R = 1 ,15835   ,522.22,454.33,406.03
XS GIS Cut Line= 3
2357236.65597196623086.8392016742357979.75205052623394.250972256
2358182.94431672623413.705997765
#Sta/Elev= 30
       0  112.63   37.13  113.17   58.12  111.76   68.46  110.29  105.79  103.46
  120.29   101.4  148.02   94.78  186.38   91.29  220.05    90.4  249.27   90.23
  289.21   88.56  333.21   88.29  352.11   89.11  397.64   88.17  418.27   88.28
  428.97   85.74  436.27   88.28  449.77   89.07  475.06   88.48  522.39   88.31
   566.6   88.98  608.97    88.7  632.45   91.06  693.37   93.58  728.71   96.31
  784.62   99.41  841.92  103.59   863.5  104.42  894.56104.5502 1008.29   106.5
#Mann= 5 ,-1 , 0
       0     .09       0  148.02     .07       0  418.27     .05       0
  436.27    .075       0  894.56     .04       0
#XS Ineff= 2 , 0
       0  304.41   94.33     550       0   94.17
Permanent Ineff=
       F       F
Bank Sta=418.27,436.27
XS Rating Curve= 0 ,0
Exp/Cntr=0.3,0.1

Type RM Length L Ch R = 1 ,15381   ,302.42,250.27,224.88
XS GIS Cut Line= 2
2356995.66043423623753.5773382042357968.69407314623664.065619811
#Sta/Elev= 30
       0  111.19   38.85  110.02  127.75  105.56  184.94  100.52  205.43   99.25
  213.58   97.91  273.33   95.23  292.39   95.12  325.53   93.43  370.83   92.64
   413.3   91.19  445.42   90.77  463.45   89.72  505.47   88.67  518.75   87.45
  531.52   87.95  556.45   87.13  607.02   86.83  611.86   85.97  617.21   84.23
  624.63   86.84  640.92   87.52     696    87.4  705.35   88.21  735.13   92.23
  764.91    95.4  875.39   99.21  912.34   98.89  933.37   99.22  977.14  100.17
#Mann= 5 ,-1 , 0
       0    .085       0  370.83     .07       0  607.02     .05       0
  624.63    .075       0  933.37     .04       0
Bank Sta=607.02,624.63
XS Rating Curve= 0 ,0
Exp/Cntr=0.3,0.1

Type RM Length L Ch R = 1 ,15130   ,487.01,482.95,459.61
BEGIN DESCRIPTION:
Surveyed Section
END DESCRIPTION:
XS GIS Cut Line= 6
2357263.02588867624179.549418181    2357575.2142     623970.7984
2357590.04310003623958.7134000212357624.45680003623945.982900009
2357682.54650003623920.2750999932357945.03437845623814.754179463
#Sta/Elev= 30
       0  102.63    34.7   98.65  104.29   94.68  131.62   93.48  180.61   93.36
  252.29   90.41  277.63   88.89  313.87   86.81  326.37   86.56     373   86.69
 394.625   86.26 420.579    86.4 421.963   86.07  433.25   84.38  444.66   83.65
  453.21   85.05 470.049   86.06 471.912   86.35  504.37   86.14  525.52   86.56
  544.97   87.72  570.98   91.72  586.92   93.07  606.61   96.66  629.51   98.07
  650.51   100.6  655.48  100.61  676.43   99.95  744.25  100.66  778.11  100.34
#Mann= 5 ,-1 , 0
       0    .085       0  277.63     .07       0 421.963     .05       0
 470.049    .075       0  655.48     .04       0
Bank Sta=421.963,470.049
XS Rating Curve= 0 ,0
Exp/Cntr=0.3,0.1

Type RM Length L Ch R = 1 ,14647   ,405.39,460.85,500.41
XS GIS Cut Line= 2
2357575.70752187 624551.142083692358228.26049545624111.575150087
#Sta/Elev= 30
       0  101.96    5.98  101.97   48.59   102.3  132.25   96.48  199.59    92.5
   246.4   88.25  258.43   88.21  281.91   86.95  287.65    86.9  323.85   86.71
  329.34   86.06  376.45   85.21   393.5   86.06  408.15   85.42  414.25   82.55
   422.8   83.56  424.11   85.21  424.93   85.42  426.28   85.74  430.63   85.83
  442.08   85.64  497.94   85.88  511.55   86.25  611.94   96.08  623.38   96.21
  646.77   97.83  659.97   97.97  695.59  100.07   719.6  101.21  786.79  100.54
#Mann= 6 ,-1 , 0
       0    .045       0    5.98     .09       0  287.65     .07       0
  408.15     .05       0  424.93    .075       0   719.6     .04       0
Bank Sta=408.15,424.93
XS Rating Curve= 0 ,0
Exp/Cntr=0.3,0.1

Type RM Length L Ch R = 1 ,14187   ,314.04,347.35,332.7
XS GIS Cut Line= 3
2357695.79539549624795.8494487852358246.69365878624721.119801164
2358389.13292992624730.140989661
#Sta/Elev= 30
       0  105.78   13.02  106.02   18.85  105.92   36.24  104.51  129.85   99.12
  136.03   98.39  188.42   86.77  204.99   85.01  206.46   84.99  247.09   84.73
  262.24   85.12   270.9   83.81  271.33   84.27  279.51   84.84   286.2   84.31
  353.38    84.5  365.95   84.02  374.17    83.6  387.41   81.33  400.74      84
  434.73   84.89  468.75   85.33  474.26    85.6  498.51   86.92  526.49   91.64
     568   97.02  615.06  100.28  641.64  101.82  655.23  102.51  698.67  104.16
#Mann= 5 ,-1 , 0
       0     .09       0  206.46     .07       0  365.95     .05       0
  400.74     .07       0  474.26    .075       0
Bank Sta=365.95,400.74
XS Rating Curve= 0 ,0
Exp/Cntr=0.3,0.1

Type RM Length L Ch R = 1 ,13839   ,244.35,268.35,241.54
XS GIS Cut Line= 3
2357537.18876992625006.5696798562357800.02260654 625083.60718368
2358348.34836906 625058.68328537
#Sta/Elev= 30
       0  103.62   70.31  101.09  117.74  100.84  155.18     100  199.12   96.29
  229.64   92.03  246.09    90.8  263.06    87.5  284.55   84.89  291.09   85.21
  323.35   85.14  338.18   84.55  360.31   85.06  376.23   84.52   392.5   84.72
  458.69   83.92  491.67   83.67  497.58   83.17  502.81   82.71  510.69   80.34
  523.51   83.18  524.65   83.57  538.15   83.92  581.95   83.32  626.88   85.96
  665.08   88.69  691.08   89.81  726.26   94.81  760.33   96.91  822.78  103.04
#Mann= 6 ,-1 , 0
       0    .045       0  117.74     .09       0  458.69     .07       0
  497.58     .05       0  523.51     .07       0  626.88     .07       0
#XS Ineff= 2 , 0
       0  350.49   88.42               0
Permanent Ineff=
       F       F
Bank Sta=497.58,523.51
XS Rating Curve= 0 ,0
Exp/Cntr=0.3,0.1

Type RM Length L Ch R = 1 ,13571   ,412.23,401,383.98
XS GIS Cut Line= 4
2357496.40420906 625369.099109652357958.62923205625319.251313031
2358264.51343843625303.3906504962358389.13292992625335.111975595
#Sta/Elev= 30
       0  101.55   49.19   99.94   64.05   99.32   79.34   99.04  154.68   96.52
  167.76   96.45  197.98   95.66  214.22   95.06  250.27   94.82  283.17   94.03
  298.37      94   329.7   93.66  386.91   92.11  398.69   91.78  407.45   91.14
  416.74   90.83  487.05   84.12  502.89 83.6593  521.55   82.78  530.64   82.53
  543.94   79.76  557.37   82.42     670    84.1   729.8   88.35  739.27    88.7
  758.63   89.65  764.11   89.64  769.22   90.41  833.02    95.2  899.79  101.09
#Mann= 6 ,-1 , 0
       0    .045       0  386.91     .09       0  502.89     .07       0
  530.64     .05       0  557.37     .07       0  739.27     .07       0
Bank Sta=530.64,557.37
XS Rating Curve= 0 ,0
Exp/Cntr=0.3,0.1

Type RM Length L Ch R = 1 ,13170   ,520.23,547.71,497.82
XS GIS Cut Line= 3
2357679.93473293625776.9447181522358057.15789197  625698.7334539
2358321.15866186625684.046551749
#Sta/Elev= 30
       0  102.31   20.62  101.74   52.56   99.56   61.79    98.9   94.12   94.65
   131.6   89.09  154.07    86.8  166.75   85.22  171.05   84.89  206.83    82.1
  215.07   81.65  219.01   82.03  234.78   81.67   278.9   81.18  296.24    81.8
  310.49   81.99  323.61   81.76  342.13   81.11  355.82    78.4  372.07   81.09
   380.4   81.42  430.89   81.41  462.46    81.7  501.14   83.99  521.51   84.47
  531.29   86.12  551.48   89.98  574.94   91.12  613.05   96.78  649.65  101.22
#Mann= 6 ,-1 , 0
       0    .085       0   52.56    .075       0  171.05     .07       0
  342.13     .05       0  372.07     .07       0  531.29     .07       0
Bank Sta=342.13,372.07
XS Rating Curve= 0 ,0
Exp/Cntr=0.3,0.1

Type RM Length L Ch R = 1 ,12622   ,856.5,914.86,873.59
XS GIS Cut Line= 3
2357650.47921677626277.6884930132357820.51717649626295.864231274
2358545.47374652626069.234070882
#Sta/Elev= 30
       0   98.33   47.07   96.97  119.48   96.02  164.26    96.5  237.52   94.11
  247.72   92.81   266.3   91.45  276.74   89.61  320.12   85.88  330.41   83.91
  358.46   81.72   398.4   80.76  431.62    80.8  440.77   81.62  468.35   81.43
  495.94   80.82   616.5   80.54  623.01   80.04  637.77   76.62  641.04   76.91
  644.39   79.46  646.37   79.97  649.35   80.74  657.26   80.75   733.4   79.72
  781.02   83.04   804.4   88.96  846.42   97.84  878.34  103.58  930.56  107.44
#Mann= 7 ,-1 , 0
       0     .11       0  247.72    .075       0  468.35     .07       0
  623.01     .05       0  646.37     .07       0  657.26     .09       0
  781.02     .07       0
#XS Ineff= 2 , 0
       0     500    86.2               0
Permanent Ineff=
       F       F
Bank Sta=623.01,646.37
XS Rating Curve= 0 ,0
Exp/Cntr=0.3,0.1

Type RM Length L Ch R = 1 ,11707   ,618.83,637,615.41
XS GIS Cut Line= 2
2357915.61578178627103.0965784942358871.02502561626915.110963404
#Sta/Elev= 30
       0  104.36   19.21  103.37   52.57  100.75   58.45   99.85   98.99   99.66
  140.18   97.45   157.1   97.33  215.32   89.73  238.87   88.07  307.32   80.72
  340.93   79.53  409.08   79.53   466.9   77.89  478.73   77.26  507.09   77.58
   517.5    77.2  529.69   74.58  534.97   76.86   540.4    77.2  553.34   78.07
  620.58   79.96  650.55   81.43   708.1   82.14   795.6   84.87  819.03   85.14
  836.11   87.96  844.71   90.28  855.19    93.1  886.34   99.18  973.73  101.13
#Mann= 5 ,-1 , 0
       0      .1       0   466.9     .07       0   517.5     .05       0
   540.4     .09       0  844.71     .04       0
Bank Sta=517.5,540.4
XS Rating Curve= 0 ,0
Exp/Cntr=0.3,0.1

Type RM Length L Ch R = 1 ,11070   ,574.36,645.48,628.84
XS GIS Cut Line= 2
2358167.08365417627691.5532691332359019.02781415627492.162082762
#Sta/Elev= 30
       0  107.44   27.08  105.75   80.18  101.75  114.02   96.24  131.69   92.07
  166.53   86.73  176.82   85.95  180.89   85.13  230.62   79.08  237.41   78.65
  264.41   78.38  278.66   77.85  291.42   76.43  351.46   76.56  365.51   76.85
   369.7   76.64  371.34   76.37  381.24   72.92  389.49   76.32  391.55   76.64
   417.6    78.1  439.37   77.71  496.12   78.03  536.98   77.73  630.12   78.69
  739.49   87.79  763.94   88.15  797.11   90.62  850.66   93.77  874.97   96.22
#Mann= 4 ,-1 , 0
       0      .1       0  264.41     .07       0   369.7     .05       0
  391.55     .07       0
Bank Sta=369.7,391.55
XS Rating Curve= 0 ,0
Exp/Cntr=0.3,0.1

Type RM Length L Ch R = 1 ,10425   ,394.65,408.83,354.75
XS GIS Cut Line= 3
2358198.80497928628244.4106495382358468.43624267628192.297043994
2359116.45759837628203.626088709
#Sta/Elev= 30
       0   94.67    30.2   93.58  113.76   88.56  157.21   86.91  227.87   80.98
   235.8   80.97   260.9   79.28  297.85   76.25  337.82   75.93  348.88   74.75
  357.48   71.15   362.5   73.55  369.85   74.75  386.81   75.72  437.67   76.89
  499.99   76.69  529.51   77.08  545.52   78.76   565.2   79.02  596.69   80.69
  632.92   80.62   640.7   79.97  665.76   80.07  711.94   84.52  733.03   85.74
  787.22   87.99   817.9   89.93  868.87   91.71  892.15   93.39  922.74   93.68
#Mann= 5 ,-1 , 0
       0      .1       0  297.85     .07       0  348.88     .05       0
  369.85     .09       0  545.52     .07       0
Bank Sta=348.88,369.85
XS Rating Curve= 0 ,0
Exp/Cntr=0.3,0.1

Type RM Length L Ch R = 1 ,10016   ,181.34,193.99,179.86
XS GIS Cut Line= 2
2358046.99578054628656.7878759212359016.76200525628498.181250378
#Sta/Elev= 30
       0   93.07   71.67   90.53   80.36   90.47  154.87   87.53  186.75   85.65
  220.39    82.4  236.82   80.35  257.59    79.2  315.35   77.33  356.18   76.43
  480.04   74.92  505.94   73.17  527.32   69.86  543.94   72.93  555.07   73.54
  577.13    74.6  641.62   75.97  673.61   76.32  684.37   76.42  700.31   77.94
  722.56   78.62  779.07   78.86  795.17   79.15  818.66   80.03  841.18   81.86
  842.64   82.27   901.1   88.14  924.79   89.76  951.26   92.26  982.65    93.1
#Mann= 4 ,-1 , 0
       0     .09       0  505.94     .05       0  555.07     .09       0
  673.61     .07       0
Bank Sta=505.94,555.07
XS Rating Curve= 0 ,0
Exp/Cntr=0.5,0.3

Type RM Length L Ch R = 1 ,9822    ,71.37,79.94,80.06
BEGIN DESCRIPTION:
Surveyed Section
END DESCRIPTION:
XS GIS Cut Line= 6
2357989.23984104 628911.286231162358315.40649298628797.386765406
2358764.26770002628722.1455000042358944.44217885628679.604363337
2359023.39521764628648.5408726782359151.53211658628582.530955017
#Sta/Elev= 30
       0   94.17    8.73   93.44   21.86   93.77   39.37   92.23   48.14   90.72
   75.71    89.3  107.01   89.28  235.12   86.41   427.2   80.53  494.98   79.75
  525.53   78.28  564.08   78.39  585.91   77.26 615.542   77.27  651.15   75.68
 666.894   75.72 672.382   73.05 691.595   68.87 699.117    69.7 703.689   71.13
 706.357   73.04  711.33   75.97  733.19   77.43 801.856   80.41  820.98   82.43
 1025.71   90.03  1093.1   94.63 1099.28   96.16 1143.41   97.17 1212.85   96.78
#Mann= 5 ,-1 , 0
       0     .09       0 672.382     .05       0 706.357     .09       0
  733.19     .07       0  1093.1    .045       0
#XS Ineff= 2 , 0
       0  667.38   80.49  710.63       0   80.99
Permanent Ineff=
       F       F
Bank Sta=672.382,706.357
XS Rating Curve= 0 ,0
Exp/Cntr=0.5,0.3

Type RM Length L Ch R = 2 ,9781    ,,,
BEGIN DESCRIPTION:
Cow Branch Road
END DESCRIPTION:
Bridge Culvert--1,0,-1,-1, 0
Deck Dist Width WeirC Skew NumUp NumDn MinLoCord MaxHiCord MaxSubmerge Is_Ogee
29.5,19.5,2.6,0, 49, 49, , , 0.98, 0, 1,1,,
       0   26.86   70.54  149.55  192.44  234.49  315.28  378.05  423.93  453.97
 488.246 544.354 602.532 661.497 690.388 726.031 782.634 840.282 899.044  910.74
  941.74  988.55 1010.94 1073.02  1082.2 1082.69 1083.04 1098.73 1103.98 1110.49
 1115.12 1125.54 1130.38  1133.3 1144.68 1147.58 1152.61 1158.68 1171.07 1171.89
 1172.83 1175.42 1184.24 1194.84    1195 1195.14 1211.85 1217.08 1222.38
   97.06    95.5   93.26   90.01    88.2   87.05   84.95   83.45   82.13    81.4
   80.98   80.71   80.49   80.69   80.72    81.2   82.52   84.76   87.02   87.44
   88.58   90.36   91.11   93.14   93.41   93.43   93.44   93.99   94.08   94.05
   94.24   94.58   94.47   94.43   94.85   94.88   95.01   95.05   95.43   95.46
   95.49   95.47   95.52   95.93   95.94   95.94   96.07    96.3   96.32
                                                                                
                                                                                
                                                                                
                                                                                
                                                                        
       0   26.86   70.54  149.55  192.44  234.49  315.28  378.05  423.93  453.97
 488.246 544.354 602.532 661.497 690.388 726.031 782.634 840.282 899.044  910.74
  941.74  988.55 1010.94 1073.02  1082.2 1082.69 1083.04 1098.73 1103.98 1110.49
 1115.12 1125.54 1130.38  1133.3 1144.68 1147.58 1152.61 1158.68 1171.07 1171.89
 1172.83 1175.42 1184.24 1194.84    1195 1195.14 1211.85 1217.08 1222.38
   97.06    95.5   93.26   90.01    88.2   87.05   84.95   83.45   82.13    81.4
   80.98   80.71   80.49   80.69   80.72    81.2   82.52   84.76   87.02   87.44
   88.58   90.36   91.11   93.14   93.41   93.43   93.44   93.99   94.08   94.05
   94.24   94.58   94.47   94.43   94.85   94.88   95.01   95.05   95.43   95.46
   95.49   95.47   95.52   95.93   95.94   95.94   96.07    96.3   96.32
                                                                                
                                                                                
                                                                                
                                                                                
                                                                        
BR Coef=-1 , 1 , 0 ,1.25, 0 ,,,0.8,0,2,0,
WSPro=,,,, 1 ,,,, 0 ,,,, 0 ,,,,-1 ,-1 ,-1 , 0 , 0 , 0 , 0 , 0
Multiple Barrel Culv=3,6.75,10.25,55,0.024,0.9,1,34,3,68.69,67.95, 2,Culvert #1  , 0 ,13.5
   682.5   679.5   695.5   692.5
Culvert Bottom n=0.024
BC Design=,, 0 ,, 0 ,,,,,,
BC Use User HTab Curves=0
BC User HTab FreeFlow(D)= 0

Type RM Length L Ch R = 1 ,9742    ,194.61,205.53,189.59
BEGIN DESCRIPTION:
Surveyed Section
END DESCRIPTION:
XS GIS Cut Line= 6
2358013.83177114628978.590460926 2358341.2927352628867.279619396
2358578.24850005628823.9244000022358670.39619999 628820.77670002
2358956.09098782 628755.968777882359185.18423146628647.246560574
#Sta/Elev= 30
       0   95.34   22.39   93.33   104.2   90.93  200.42   86.53  247.44   83.82
  321.25   82.19  402.72   79.33  452.24   76.74  531.16   78.23  546.33   77.65
  561.53   78.55  584.49   77.05 586.934   76.37  626.84   77.45 664.311   76.84
 671.574   72.92  680.05    68.1  695.01   67.89 700.805   73.16 709.532   78.86
 758.788   79.55  789.39  81.371  816.18   83.08  840.91   84.24  886.04   84.49
  967.93      89 1004.07   89.83 1019.87   89.99 1138.55    95.4 1228.82      98
#Mann= 9 ,-1 , 0
       0     .04       0   54.19    .035       0   104.2     .04       0
  200.42    .085       0 671.574     .05       0 700.805     .07       0
  789.39    .035       0  816.18     .07       0 1004.07    .035       0
#XS Ineff= 2 , 0
       0  664.38    74.7  707.63       0    74.7
Permanent Ineff=
       F       F
Bank Sta=671.574,700.805
XS Rating Curve= 0 ,0
Exp/Cntr=0.5,0.3

Type RM Length L Ch R = 1 ,9537    ,494.71,524.03,433.64
XS GIS Cut Line= 4
2358242.93191165629091.3209076822358623.32633275629007.280279741
2358656.50026485629011.703470677  2358999.297563 628956.41358389
#Sta/Elev= 30
       0   92.46   27.44   92.37   56.61   90.99   85.25   87.61  136.95   78.56
  152.69    75.8  167.65   74.87  298.15    73.7  362.17   76.15  392.91   73.82
  394.97   73.63     400   70.42  408.55   67.37  418.05   70.54  421.75   73.48
  423.04   73.82  441.28   75.34  455.31   75.13  503.96   75.72   528.4   77.38
  544.52   79.04  593.02   79.88  637.82   83.28  673.74   85.33  679.41    86.1
  706.75   87.54  712.65   88.79  721.95    91.6  744.19   92.63  770.26    94.7
#Mann= 4 ,-1 , 0
       0     .04       0  136.95    .085       0  392.91     .05       0
  423.04     .07       0
#XS Ineff= 2 , 0
       0   359.8   79.61               0
Permanent Ineff=
       F       F
Bank Sta=392.91,423.04
XS Rating Curve= 0 ,0
Exp/Cntr=0.3,0.1

Type RM Length L Ch R = 1 ,9012    ,327.69,382.46,345.5
XS GIS Cut Line= 2
 2358307.5638082629646.9463809882359025.82524098629354.657028213
#Sta/Elev= 30
       0   90.36   34.88   89.13   45.38   88.24  105.69   85.93  137.42   84.23
  174.29   84.62  193.19   83.86  196.54   84.05  226.73   83.31  254.48    83.1
  263.09   82.22  320.01   78.57  330.32   79.02  338.25   78.45  342.75   78.13
  366.14   74.66  435.53   72.31  461.82      73   528.1   73.65  619.51    73.4
  623.29   73.12  643.23   66.44  653.68   72.15  659.75   73.18  663.05   73.55
  664.99    75.2  684.19   79.93  722.19   85.14  751.25   90.21  775.46   92.83
#Mann= 5 ,-1 , 0
       0     .04       0  338.25    .085       0  623.29     .05       0
  659.75     .09       0  684.19     .07       0
Bank Sta=623.29,659.75
XS Rating Curve= 0 ,0
Exp/Cntr=0.3,0.1

Type RM Length L Ch R = 1 ,8630    ,452.62,488.88,466.15
XS GIS Cut Line= 4
2358525.08146609629884.8563192642358687.46260148629832.205390722
 2359039.1062815 629717.202426212359134.58406991629676.401897162
#Sta/Elev= 30
       0   90.75   21.67   89.05   49.23   86.54   63.35   84.61   71.01   83.56
   89.32   82.59  125.64   79.77  144.94   78.83  154.56   77.73  173.44   76.47
  185.94   75.51  218.76   73.54  298.25   72.75  303.79   72.49  357.68   72.44
  364.56   71.92  367.34   71.71  369.12   71.23  386.58   65.63  395.72   69.96
  402.38   71.46  406.15   71.73  408.75   71.92  443.19   73.42  456.33   72.77
  473.81   72.69  520.45    73.2  548.35   77.34  633.48   88.92  644.51   90.25
#Mann= 6 ,-1 , 0
       0     .04       0   63.35      .1       0  173.44    .085       0
  364.56     .05       0  408.75     .09       0  548.35     .07       0
Bank Sta=364.56,406.15
XS Rating Curve= 0 ,0
Exp/Cntr=0.3,0.1

Type RM Length L Ch R = 1 ,8141    ,160.93,217.35,172.28
XS GIS Cut Line= 3
2358661.03000227630315.3600171212359337.67167017630093.173656404
2359374.75981714630070.652652025
#Sta/Elev= 30
       0   91.33   57.88   89.46   94.97   88.53  121.82   85.71  158.69   80.92
   189.1   78.66  200.59   78.39  219.44   77.41  257.71    76.5   334.2   72.15
  396.81   70.99  404.15   70.63  411.03   69.85  446.17   70.43  455.98   70.03
  467.23   70.13  471.26   69.44  483.61   64.71  493.11   68.63  496.05   70.18
  530.46   70.39  568.79   71.87  601.29    71.5  645.72   71.71  680.61   73.08
  702.57   72.99  716.89   74.64  723.52   76.21  728.86   76.62  755.58   81.74
#Mann= 5 ,-1 , 0
       0    .045       0   57.88      .1       0  467.23     .05       0
  496.05     .09       0  645.72     .07       0
#XS Ineff= 2 , 0
       0                  681.37       0   76.68
Permanent Ineff=
       F       F
Bank Sta=467.23,496.05
XS Rating Curve= 0 ,0
Exp/Cntr=0.3,0.1

Type RM Length L Ch R = 1 ,7924    ,544.37,631.64,573.74
XS GIS Cut Line= 3
2358679.15647374630462.6375979632359331.03688377630281.159271523
2359426.87342262630245.119940102
#Sta/Elev= 30
       0   90.62   46.35   89.29      93   88.11  134.34   86.08  189.85   81.81
   236.8   80.72  270.27   78.13  287.07   78.55  322.67   76.24  362.79   71.66
  372.89   71.48  381.28   71.88  393.15   70.45   408.5   69.51  413.64   69.18
   417.1   65.58   422.8   64.38  429.04   69.15  434.97   69.49  444.92   70.07
  492.34   70.04   501.3   69.68  518.85      70  540.02   69.12  576.61    70.2
  673.18    71.1  693.13   73.66  736.47   79.32  751.02   80.22  779.06   83.42
#Mann= 5 ,-1 , 0
       0    .045       0   46.35      .1       0   408.5     .05       0
  434.97     .09       0  693.13     .07       0
Bank Sta=408.5,434.97
XS Rating Curve= 0 ,0
Exp/Cntr=0.3,0.1

Type RM Length L Ch R = 1 ,7292    ,516.67,545.02,534.54
XS GIS Cut Line= 3
2358717.67522565630870.4832064662358971.44582653 630920.33100307
2359527.86888075 630840.69292587
#Sta/Elev= 30
       0   88.57   12.57   87.65   46.02   86.11   54.62   85.32   96.75   82.56
  137.81   82.51  174.36   81.76  193.19   81.79  238.56   81.16  257.68   80.61
  340.26   75.06  357.09   73.44  394.07   70.22   425.3   69.26  435.68   69.03
  462.12    69.1  509.48   68.44  540.74   68.85   554.9   68.23  570.07    63.5
  582.68   68.22  596.97   69.09   613.5   70.68  650.95   73.15  684.21   74.96
  715.67   78.46  724.88   79.08  739.33   80.53  780.21    89.1  820.71   90.61
#Mann= 4 ,-1 , 0
       0     .04       0  357.09      .1       0   554.9     .05       0
  582.68     .09       0
Bank Sta=554.9,582.68
XS Rating Curve= 0 ,0
Exp/Cntr=0.3,0.1

Type RM Length L Ch R = 1 ,6747    ,268.72,330.38,272.55
XS GIS Cut Line= 3
2358700.73217428631362.6294572352358892.14251371631425.606395811
2359567.35357668631389.353452832
#Sta/Elev= 30
       0   90.02   22.58   88.91   91.07   87.67  140.48   87.13  174.98   86.09
  195.45   86.05  219.21   85.23  252.52    82.4  280.61   80.79  346.95   76.17
  399.63   71.09  425.61   68.98  443.09   69.16   487.2    68.9  543.19   67.22
  551.64   66.76  570.07   62.62  585.43   67.22  592.93    67.6   593.1   68.94
  646.27   69.54  680.72   70.86  712.96   76.52  730.11   78.67   734.2   79.68
  773.64   84.36  794.99   85.08  826.85   86.89  861.26   89.22  877.69   90.78
#Mann= 3 , 0 , 0
       0      .1       0  543.19     .05       0  585.43     .09       0
Bank Sta=543.19,585.43
XS Rating Curve= 0 ,0
Exp/Cntr=0.3,0.1

Type RM Length L Ch R = 1 ,6417    ,306.8,384.95,319.72
XS GIS Cut Line= 2
2358710.87779887631713.3641307062359512.97416222631654.453098357
#Sta/Elev= 30
       0    88.2   49.14   85.74   88.23   84.17   94.76   84.35  107.29    84.1
  134.07   82.74   176.8   78.85  233.24   74.83  254.69   72.04  289.62   71.17
  336.36   70.42  352.16    69.5  422.21   67.67  465.09   68.49  482.77   67.72
  535.83   67.33   568.7   66.32  592.01   66.79  629.81   66.57  653.05   67.14
  668.36   67.27  672.18   67.07  690.02   62.02  703.56   67.09  704.71   67.27
  708.71   69.22  713.56   70.12  718.27   71.99  793.73   85.79  804.26   88.35
#Mann= 3 , 0 , 0
       0      .1       0  672.18     .05       0  703.56     .09       0
Bank Sta=672.18,703.56
XS Rating Curve= 0 ,0
Exp/Cntr=0.3,0.1

Type RM Length L Ch R = 1 ,6032    ,507,667.4,504.92
XS GIS Cut Line= 2
2358806.04177418632012.4509102552359503.91092648631962.603113666
#Sta/Elev= 30
       0   91.43   34.19   89.81   42.83   89.74    59.1   88.38   69.34   87.69
   79.24   86.71  115.83   83.82  147.69   80.46  169.38   78.93  207.66   73.71
  218.82   72.51  228.68   71.16  232.72      71  261.77    70.5  310.28   69.09
  319.36   68.68  355.07   66.54  378.21   65.72  398.58   65.73  498.23   67.09
  507.02   66.74  530.64   66.35  547.86   61.21  563.56   66.35  570.63   67.37
  583.26   68.53  594.73   69.47  641.98    76.3  695.92   88.67  699.65   89.13
#Mann= 3 , 0 , 0
       0      .1       0  530.64     .05       0  563.56     .09       0
Bank Sta=530.64,563.56
XS Rating Curve= 0 ,0
Exp/Cntr=0.3,0.1

Type RM Length L Ch R = 1 ,5364    ,357.34,493.26,358.75
XS GIS Cut Line= 4
2358731.69451089632470.6387886112358901.98736222632503.812720686
2359545.56164452632461.7924067232359744.60523699632395.444542572
#Sta/Elev= 30
       0   89.81   16.32   89.47   44.14   90.16   95.17   87.52  102.57   87.76
  131.95   86.41  176.16   85.65  220.79   83.64  261.57   80.34   281.6   79.84
   391.2   69.64   431.1   69.02  457.41   67.08  520.78   65.17  530.17   63.43
  542.99    60.2  555.82   63.77  563.65   65.26  631.22   65.44  683.62   66.81
  738.48   67.26  813.76   76.33  836.19   77.46  864.17   80.37  919.57   81.62
  929.48   82.47  942.65   82.69  990.38   86.09 1013.55   86.24 1028.25   86.52
#Mann= 4 ,-1 , 0
       0      .1       0  520.78     .05       0  563.65    .075       0
 1013.55    .032       0
Bank Sta=520.78,563.65
XS Rating Curve= 0 ,0
Exp/Cntr=0.3,0.1

Type RM Length L Ch R = 1 ,4871    ,570.4,636.77,572.31
XS GIS Cut Line= 4
2358830.96567248632909.7112489492359176.22520073632820.070873156
2359523.44568978632806.8013003322359703.30211285632819.078891531
#Sta/Elev= 30
       0   89.29   32.72    87.7   99.12   84.01  138.88   79.88   159.6   78.81
   186.8   75.39  251.78   69.62  259.64   68.76  304.87   67.59   342.4    64.5
  358.07   63.69  367.27   63.74  385.63   62.57  402.61   59.44  419.99   62.53
  448.49   63.98  477.78   62.07   526.7   64.83  544.66   65.01  558.35   64.65
  590.45   64.35  649.56   69.41  693.31   74.31  722.76   76.92  757.12   79.07
  798.58   82.52  812.16   83.29  840.05    85.6  847.56   86.49  884.46   88.08
#Mann= 4 ,-1 , 0
       0    .045       0   32.72      .1       0  385.63     .05       0
  419.99     .09       0
Bank Sta=385.63,419.99
XS Rating Curve= 0 ,0
Exp/Cntr=0.3,0.1

Type RM Length L Ch R = 1 ,4234    ,639.6,755.14,648.22
XS GIS Cut Line= 2
2358776.58625802633371.9362719212359857.37712049 633390.06274341
#Sta/Elev= 30
       0   83.97   54.05   81.19   87.21   80.66  110.33   77.65  140.94      76
     195   74.36  227.18   72.44  282.53   66.84  329.42   66.13  356.52    64.5
  385.65   64.95  392.32   64.56   455.5   64.52  485.67    62.2  529.33   62.99
  568.65   61.33  573.55   59.32  590.02   57.62     608   60.26  614.23   60.66
  633.47   60.87  692.46   63.56  728.49   62.86  831.74   69.15   877.6   70.68
  912.55   73.02  929.04    73.1 1016.46   78.85 1060.76   84.09 1080.94   86.01
#Mann= 5 ,-1 , 0
       0    .045       0   54.05     .07       0     195      .1       0
  568.65     .05       0  614.23     .09       0
#XS Ineff= 2 , 0
       0  310.29   68.42               0
Permanent Ineff=
       F       F
Bank Sta=568.65,614.23
XS Rating Curve= 0 ,0
Exp/Cntr=0.3,0.1
