--- Black_Creek_US_FINAL.prj (project) ---

Proj Title=Black Creek US
Current Plan=p02
Default Exp/Contr=0.3,0.1
English Units
Geom File=g01
Flow File=f01
Flow File=f02
Plan File=p01
Plan File=p02
Y Axis Title=Elevation
X Axis Title(PF)=Main Channel Distance
X Axis Title(XS)=Station
BEGIN DESCRIPTION:
NEUSE RIVER BASIN
Little Contentnea Creek Sub-basin
BLACK CREEK 1
(Flood Hazard, Floodway) Model
Prepared by: Andrew J. Bonner   Date: 11/21/2002
Watershed Concepts
3333 Regency Pkwy
Cary, North Carolina 27511
END DESCRIPTION:
DSS Export Rating Curves= 0
DSS Export Rating Curve Sorted= 0
DSS Export Volume Flow Curves= 0
DXF OffsetX= 0
DXF OffsetY= 0
DXF ScaleX= 1
DXF ScaleY= 10

--- Black_Creek_US_FINAL.p02 (plan) ---

Plan Title=Multi_Profile
Program Version=4.00
Short Identifier=Multi_Profile
Geom File=g01
Flow File=f02
Subcritical Flow
K Sum by GR= 0
Std Step Tol= 0.01
Critical Tol= 0.01
Num of Std Step Trials= 20
Max Error Tol= 0.3
Flow Tol Ratio= 0.001
Split Flow NTrial= 30
Split Flow Tol= 0.02
Split Flow Ratio= 0.02
Log Output Level= 0
Friction Slope Method= 1
Unsteady Friction Slope Method= 2
Unsteady Bridges Friction Slope Method= 1
Parabolic Critical Depth
Global Vel Dist= 0 , 0 , 0
Global Log Level= 0
CheckData=True
Encroach Param=-1 ,10,10, 2
Computation Interval=1HOUR
Output Interval=1HOUR
Run HTab= 0
Run UNet= 0
Run PostProcess= 0
Run WQNet= 0
UNET Theta= 1
UNET Theta Warmup= 1
UNET ZTol= 0.02
UNET ZSATol= 0.1
UNET MxIter= 20
UNET MaxInSteps= 20
UNET DtIC= 0
UNET DtMin= 0
UNET MaxCRTS= 20
UNET WFStab= 2
UNET SFStab= 1
UNET WFX= 1
UNET SFX= 1
UNET DSS MLevel= 4
UNET DZMax Abort= 100
UNET Convert EG Bridges=-1
UNET Use Existing IB Tables=-1
UNET Froude Reduction=False
UNET Froude Limit= 1
UNET Froude Power= 10
UNET Time Slicing=0,0, 5
Instantaneous Interval=1HOUR
Write IC File= 0
Echo Input=False
Echo Output=False
Write Detailed= 0
Detailed Automatic Start=False, 10
WQ ULTIMATE=-1
WQ Max Comp Step=1HOUR
WQ Output Interval=15MIN
WQ Output Selected Increments= 0
WQ Output face flow=0
WQ Output face velocity=0
WQ Output face area=0
WQ Output face dispersion=0
WQ Output cell volume=0
WQ Output cell surface area=0
WQ Output cell continuity=0
WQ Output face conc=0
WQ Output face dconc_dx=0
WQ Output face courant=0
WQ Output face peclet=0
WQ Output face adv mass=0
WQ Output face disp mass=0
WQ Output cell mass=0
WQ Output cell source sink temp=0
WQ Output cell source sink nsm=0
WQ Output MaxMinRange=-1
WQ Daily Max Min Mean=-1
WQ Daily Range=0
WQ Daily Time=0
WQ Create Restart=0
WQ Fixed Restart=0
WQ System Summary=False
Sorting and Armoring Iterations= 10
XS Update Threshold= 0.02
Hydraulics Update Threshold= 0.02
Energy Slope Method= 1
Volume Change Method= 0
XS Weighting Method= 0
Number of US Weighted Cross Sections= 1
Number of DS Weighted Cross Sections= 1
Upstream XS Weight=0.25
Main XS Weight=0.5
Downstream XS Weight=0.25
Number of DS XS's Weighted with US Boundary= 1
Upstream Boundary Weight= 1
Weight of XSs Associated with US Boundary= 0
Number of US XS's Weighted with DS Boundary= 1
Downstream Boundary Weight= 0.5
Weight of XSs Associated with DS Boundary= 0.5
Sediment Output Level= 4
Mass or Volume Output= 0
Output Increment Type= 1
Profile and TS Output Increment= 10
XS Output Flag= 0
XS Output Increment= 10
Disregard all LS=0
Disregard all Conn=0
Disregard all Breaches=0
Disregard all Pumps=0

--- Black_Creek_US_FINAL.p01 (plan) ---

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Plan Title=100 Year Single
Short Identifier=Plan01
Geom File=g01
Flow File=f01
Encroach River=Black Ck US
Encroach Reach=Reach - 1
Encroach Node=84618.4
       4      .7
Encroach Node=84145.9
       4      .7
Encroach Node=83545.1
       4      .7
Encroach Node=83073.7
       4      .7
Encroach Node=82395.0
       4      .7
Encroach Node=81771.0
       1    4815    5203
Encroach Node=81650.1
       1    4940    5203
Encroach Node=81606.1
       1    4940    5203
Encroach Node=81208.6
       4      .7
Encroach Node=80730.4
       4      .7
Encroach Node=79961.2
       4      .7
Encroach Node=79175.8
       4      .7
Encroach Node=78528.0
       4      .7
Encroach Node=77759.0
       4      .7
Encroach Node=76971.5
       4      .7
Encroach Node=76392.7
       4      .7
Encroach Node=75721.6
       1    4850    5200
Encroach Node=74999.3
       1    4825    5125
Encroach Node=74467.7
       1    4600    5030
Encroach Node=73750.6
       4      .7
Encroach Node=73286.3
       4      .7
Encroach Node=73241.3
       4      .7
Encroach Node=72732.8
       4      .7
Encroach Node=72169.2
       4      .7
Encroach Node=71638.5
       4      .7
Encroach Node=71148.2
       4      .7
Encroach Node=70684.9
       4      .7
Encroach Node=70247.2
       4      .7
Encroach Node=69332.9
       1    4500    5250
Encroach Node=68725.6
       1    4600    5300
Encroach Node=68090.4
       1    4600    5300
Encroach Node=67467.7
       4      .7
Encroach Node=66679.7
       4      .7
Encroach Node=66140.7
       4      .7
Encroach Node=65670.2
       1    4900    5400
Encroach Node=65626.2
       1    4900    5400
Encroach Node=65043.1
       4      .7
Encroach Node=64391.3
       1    4700    5200
Encroach Node=63191.1
       1    4500    5350
Encroach Node=61980.8
       1    4700    5400
Encroach Node=60797.5
       4      .7
Encroach Node=60077.1
       4      .7
Encroach Node=59093.6
       1    4800    5150
Encroach Node=58157.0
       1    4500    5050
Encroach Node=57357.2
       4      .7
Encroach Node=56215.9
       1    4875    5375
Encroach Node=55330.0
       1    4750    5600
Encroach Node=54724.8
       4      .7
Encroach Node=54010.6
       1    4600    5100
Encroach Node=53158.6
       1    4800    5450
Encroach Node=52361.1
       4      .7
Encroach Node=51505.4
       1    4875    5394

--- Black_Creek_US_FINAL.f02 (steady flow) ---

Flow Title=Multi_Profile
Program Version=4.00
Number of Profiles= 7
Profile Names=10yr,25yr,50yr,500yr,100yr-10%,100yr-20%,100yr-35%
River Rch & RM=Black Ck US,Reach - 1       ,84618.4
     630     883    1106    2070    1505    1929    2357
River Rch & RM=Black Ck US,Reach - 1       ,83545.1
    1107    1530    1901    3469    2496    3199    3908
River Rch & RM=Black Ck US,Reach - 1       ,79175.8
    1171    1616    2005    3650    2623    3362    4108
River Rch & RM=Black Ck US,Reach - 1       ,77759.0
    1234    1701    2109    3830    2750    3525    4307
River Rch & RM=Black Ck US,Reach - 1       ,74999.3
    1343    1846    2286    4137    2965    3801    4644
River Rch & RM=Black Ck US,Reach - 1       ,73286.3
    1442    1979    2448    4414    3161    4051    4949
River Rch & RM=Black Ck US,Reach - 1       ,66679.7
    2561    3464    4248    7463    5288    6777    8281
River Rch & RM=Black Ck US,Reach - 1       ,63191.1
    2610    3529    4326    7595    5380    6895    8424
River Rch & RM=Black Ck US,Reach - 1       ,58157.0
    2826    3813    4669    8168    5777    7404    9046
River Rch & RM=Black Ck US,Reach - 1       ,54010.6
    2944    3967    4855    8477    5991    7679    9382
Boundary for River Rch & Prof#=Black Ck US,Reach - 1       , 1
Up Type= 0
Dn Type= 1
Dn Known WS=90.97
Boundary for River Rch & Prof#=Black Ck US,Reach - 1       , 2
Up Type= 0
Dn Type= 1
Dn Known WS=91.69
Boundary for River Rch & Prof#=Black Ck US,Reach - 1       , 3
Up Type= 0
Dn Type= 1
Dn Known WS=92.26
Boundary for River Rch & Prof#=Black Ck US,Reach - 1       , 4
Up Type= 0
Dn Type= 1
Dn Known WS=94.66
Boundary for River Rch & Prof#=Black Ck US,Reach - 1       , 5
Up Type= 0
Dn Type= 1
Dn Known WS=92.97
Boundary for River Rch & Prof#=Black Ck US,Reach - 1       , 6
Up Type= 0
Dn Type= 1
Dn Known WS=94.27
Boundary for River Rch & Prof#=Black Ck US,Reach - 1       , 7
Up Type= 0
Dn Type= 1
Dn Known WS=95.33
DSS Import GetInterval= 0
DSS Import GetPeak= 0
DSS Import FillOption= 0

--- Black_Creek_US_FINAL.f01 (steady flow) ---

Flow Title= 100 Year Single
Program Version=4.00
Number of Profiles= 2
Profile Names=100-Year,AFW
River Rch & RM=Black Ck US,Reach - 1       ,84618.4
    1355    1355
River Rch & RM=Black Ck US,Reach - 1       ,83545.1
    2310    2310
River Rch & RM=Black Ck US,Reach - 1       ,79175.8
    2435    2435
River Rch & RM=Black Ck US,Reach - 1       ,77759
    2559    2559
River Rch & RM=Black Ck US,Reach - 1       ,74999.3
    2771    2771
River Rch & RM=Black Ck US,Reach - 1       ,73286.3
    2963    2963
River Rch & RM=Black Ck US,Reach - 1       ,66679.7
    5097    5097
River Rch & RM=Black Ck US,Reach - 1       ,63191.1
    5190    5190
River Rch & RM=Black Ck US,Reach - 1       ,58157
    5595    5595
River Rch & RM=Black Ck US,Reach - 1       ,54010.6
    5814    5814
River Rch & RM=Black Ck US,Reach - 1       ,51505.4
    5814    5814
Boundary for River Rch & Prof#=Black Ck US,Reach - 1       , 1
Up Type= 0
Dn Type= 1
Dn Known WS=92.88
Boundary for River Rch & Prof#=Black Ck US,Reach - 1       , 2
Up Type= 0
Dn Type= 1
Dn Known WS=93.85
DSS Import GetInterval= 0
DSS Import GetPeak= 0
DSS Import FillOption= 0

--- Black_Creek_US_FINAL.g01 (geometry) ---

Geom Title=Geom 01 by CodeH2 for Windows
Program Version=4.00

River Reach=Black Ck US     ,Reach - 1
Reach XY= 30
       0.0595906       0.1092972       0.0711231       0.0767576
       0.1070924       0.0591911       0.1435229       0.0726557
       0.1772387       0.1099547       0.2095972       0.1173385
       0.2411411       0.1401956       0.3369678       0.1247765
       0.3917489       0.1603925       0.4333372       0.1606641
       0.4586376        0.200569       0.5325299       0.2309188
       0.5589706       0.2678378       0.6144675       0.2647167
       0.6297808       0.2549906       0.6509573       0.1986347
       0.6673056        0.206981       0.6806873        0.237332
       0.7011054       0.2253985       0.7414581       0.2328481
       0.7480111       0.2201559       0.7875183       0.2089576
       0.7981933       0.1978492       0.8301645       0.2159479
       0.8386719       0.2060859       0.8607269       0.2276528
       0.8630567       0.2558308         0.88121       0.2837376
       0.8790967       0.3076347       0.9264807       0.3364563

Type RM Length L Ch R = 1 ,84618.4 ,472.5,472.5,472.5
BEGIN DESCRIPTION:
Black Creek 165.0
END DESCRIPTION:
#Sta/Elev= 28
  4686.3  137.71  4696.3  136.58  4716.3  135.96  4736.3  134.31  4826.3  132.83
  4846.3  130.37  4866.3  129.07  4886.3  128.31  4906.3  127.22  4916.3  127.14
  4936.3  126.94  4996.3  127.32  4996.6  123.41  5003.4  123.41  5004.4  127.44
  5014.4  127.55  5024.4  127.13  5074.4  127.18  5094.4  126.69  5134.4  127.61
  5144.4  128.62  5164.4  129.84  5174.4  131.99  5184.4  133.59  5194.4  134.14
  5234.4  138.81  5254.4  140.09  5254.9  140.11
#Mann= 3 , 1 , 0
  4686.3     .14       0  4996.3    .048       0  5004.4     .14       0
Bank Sta=4996.3,5004.4
XS Rating Curve= 0 ,0
Exp/Cntr=0.3,0.1

Type RM Length L Ch R = 1 ,84145.9 ,600.8,600.8,600.8
BEGIN DESCRIPTION:
Black Creek 164.0
END DESCRIPTION:
#Sta/Elev= 30
  4590.5  138.53  4640.5  135.91  4660.5  133.37  4700.5   131.3  4710.5  128.64
  4720.5  127.44  4740.5  126.75  4760.5  128.13  4770.5  127.42  4780.5  125.96
  4820.5  126.96  4840.5  126.44  4860.5  126.66  4910.5  125.93  4970.5  126.04
  4993.6  125.51  4996.4  124.56  4996.6  121.56  5003.4  121.56  5003.7  124.56
  5023.6  126.22  5043.6  125.87  5073.6  126.53  5093.6  127.71  5103.6   127.9
  5113.6  128.86  5133.6  131.98  5153.6  135.72  5163.6  137.25  5201.1  140.54
#Mann= 3 , 1 , 0
  4590.5     .14       0  4996.4    .048       0  5003.7     .14       0
Bank Sta=4996.4,5003.7
XS Rating Curve= 0 ,0
Exp/Cntr=0.3,0.1

Type RM Length L Ch R = 1 ,83545.1 ,471.4,471.4,471.4
BEGIN DESCRIPTION:
Black Creek US 163.0
END DESCRIPTION:
#Sta/Elev= 30
  4403.8  137.05  4503.8   135.9  4613.8  133.84  4673.8  131.65  4743.8  130.39
  4753.8  130.02  4773.8   126.3  4793.8  125.93  4823.8  126.54  4853.8  127.95
  4864.9  127.94  4873.8  127.94  4923.8  125.55  4933.8  125.78  4943.8  125.11
  4983.8  126.41 4988.45  123.56 4991.45  120.56 5008.55  120.56 5011.55  123.56
  5030.6  126.22  5050.6  125.49  5070.6  126.31  5120.6  125.43  5160.6  125.43
  5170.8  126.61  5230.8  129.37  5270.8  133.25  5300.8  138.44    5318  139.29
#Mann= 4 , 1 , 0
  4403.8      10       0  4864.9     .14       0 4988.45    .048       0
 5011.55     .14       0
Bank Sta=4988.45,5011.55
XS Rating Curve= 0 ,0
Exp/Cntr=0.3,0.1

Type RM Length L Ch R = 1 ,83073.7 ,678.7,678.7,678.7
BEGIN DESCRIPTION:
Black Creek US 162.5
END DESCRIPTION:
#Sta/Elev= 25
  4205.2  136.16  4265.2  136.14  4305.2  133.93  4325.2  134.28  4425.2  133.06
  4435.2  133.16  4455.2  132.04  4495.2   131.7  4565.2  129.08  4585.2  127.82
  4685.2  125.02  4715.2  125.31  4735.2  124.77  4815.2  124.69  4835.2  124.25
  4855.2  124.76  4984.6  122.69  4988.6  119.69  5011.4  119.69  5015.4  122.69
  5101.5  124.22  5111.5  124.83  5161.5  135.77  5181.5  136.45  5261.2  141.92
#Mann= 3 , 1 , 0
  4205.2     .14       0  4984.6    .048       0  5015.4     .14       0
Bank Sta=4984.6,5015.4
XS Rating Curve= 0 ,0
Exp/Cntr=0.3,0.1

Type RM Length L Ch R = 1 ,82395.0 ,624,624,624
BEGIN DESCRIPTION:
Black Creek US 162.0
END DESCRIPTION:
#Sta/Elev= 24
  4300.8  131.26  4330.8  130.86  4350.8   129.8  4380.8  130.35  4560.8  124.33
  4630.8  124.35  4670.8  123.65  4720.8  124.37  4780.8  123.34  4840.8  124.22
  4850.8  123.88  4870.8  121.49  4880.8  121.36  4971.5  119.41    5028  119.41
  5045.6  122.04  5055.6  122.39  5085.6  125.16  5155.6  126.23  5205.6  130.49
  5215.6  131.71  5225.6  131.72  5245.6  132.79  5273.7  132.51
#Mann= 3 , 1 , 0
  4300.8     .14       0  4880.8    .048       0  5045.6     .14       0
Bank Sta=4880.8,5045.6
XS Rating Curve= 0 ,0
Exp/Cntr=0.5,0.3

Type RM Length L Ch R = 1 ,81771.0 ,120.9,120.9,120.9
BEGIN DESCRIPTION:
Upstream Section of Bridge/Culvert/Weir
END DESCRIPTION:
#Sta/Elev= 18
  4652.8  129.69  4692.8  128.38  4722.8  128.14  4732.8  128.35  4772.8  124.71
  4782.8  124.29  4822.8  124.03  4832.8  122.33  4842.8  119.66  4992.8  118.66
  5008.7  118.66  5168.7  119.66  5188.7  120.21  5198.7  123.35  5208.7  127.12
  5218.7  127.91  5238.7  127.37  5264.3  127.41
#Mann= 3 , 1 , 0
  4652.8     .14       0  4822.8    .048       0  5198.7     .14       0
#XS Ineff= 2 , 0
       0  4812.8  127.65  5208.7       0  127.38
Permanent Ineff=
       F       F
Bank Sta=4822.8,5198.7
XS Rating Curve= 0 ,0
Exp/Cntr=0.5,0.3

Type RM Length L Ch R = 5 ,81756.0 ,,,
BEGIN DESCRIPTION:
Newsom Millpond Dam-TOR
Structure ID: Newsom Millpond Dam
Approximate Survey Structure
END DESCRIPTION:
IW Pilot Flow=0
#Inline Weir SE= 16
  4652.8  129.68  4692.8  128.37  4722.8  128.13  4732.8  128.35  4772.8  127.84
  4909.8  127.33  4959.8  123.65  4969.8  122.35  5021.2  122.23  5031.2  123.47
  5116.5  127.24  5124.3  127.36  5208.7  127.38  5218.7  127.91  5238.7  127.39
  5264.3   127.4
IW Dist,WD,Coef,Skew,MaxSub,Min_El,Is_Ogee,SpillHt,DesHd
10,10,3,0,0.95,, 0 ,,,2,2,

Type RM Length L Ch R = 1 ,81650.1 ,44,44,44
BEGIN DESCRIPTION:
Upstream Section of Bridge/Culvert/Weir
END DESCRIPTION:
#Sta/Elev= 30
  4596.3  130.09  4821.2  124.85  4871.2  123.44  4891.2  121.94  4931.2   120.9
  4941.2  121.32  4951.2  120.27  4971.2  116.74  4981.2  115.53  4981.5  114.94
    4988  113.64    5012  113.64  5018.5  114.94  5024.2  116.43  5034.2  117.85
  5074.2  120.86  5094.2  120.82  5124.2  116.97  5144.2  117.28  5154.2  118.66
  5164.2  118.91  5174.2  118.53  5191.9  119.15  5241.9  119.21  5301.9   120.1
  5311.9  120.87  5341.9  120.85  5411.9  123.23  5431.9  122.95  5547.6  126.67
#Mann= 3 , 1 , 0
  4596.3     .14       0  4981.5    .048       0  5018.5     .14       0
#XS Ineff= 2 , 0
       0    4963   121.1    5037       0   120.8
Permanent Ineff=
       F       F
Bank Sta=4981.5,5018.5
XS Rating Curve= 0 ,0
Exp/Cntr=0.5,0.3

Type RM Length L Ch R = 3 ,81628.1 ,,,
BEGIN DESCRIPTION:
Upper BC Church Rd-TOR
Structure ID: Upper BC Church Rd
Approximate Survey Structure
END DESCRIPTION:
Bridge Culvert--1,0,-1,-1, 0
Deck Dist Width WeirC Skew NumUp NumDn MinLoCord MaxHiCord MaxSubmerge Is_Ogee
10,24,2.6,0, 53, 53, , , 0.95, 0, 1,1,,
  4596.3  4726.3  4821.2  4871.2  4875.6  4891.2  4931.2  4941.2  4951.2  4965.6
  4971.2 4972.91    4973 5026.89    5027  5034.2  5054.2  5074.2  5094.2  5124.2
  5144.2  5154.2  5164.2  5174.2  5184.2  5191.9  5211.9  5231.9  5239.9  5241.9
  5271.9  5281.9  5291.9  5301.9  5309.9  5311.9    5317  5321.9  5331.9  5341.9
    5347  5351.9  5361.9    5367  5371.9  5411.9    5427  5431.9  5441.9  5442.7
    5507    5527  5547.6
  130.15  126.86  124.91   123.5  123.17  122.24  121.61  121.45   121.3  121.07
  121.07  121.07  121.07  121.05  121.05  121.05  121.05  121.04  121.03  121.03
  121.02  121.02  121.01  121.01     121  120.97  120.91  120.85  120.82  120.84
   121.1  121.21  121.31  121.43  121.57  121.54  121.45  121.57  121.82  122.06
  122.19  122.49  123.09   123.4  123.55  124.75  125.21  125.29  125.48  125.49
  126.79  126.17  126.73
  130.15  126.86  124.91   123.5  123.17     122  120.96  121.38  120.33  117.79
   116.8  116.59  119.59  119.57  116.89  117.91  119.07  120.92  120.88  117.03
  117.34  118.72  118.97  118.59  118.77  119.21  119.15  119.54  119.32  119.27
  119.99  119.82  120.32  120.16  120.78  120.93  120.75  120.58  121.04  120.91
  121.23  121.53  121.39  121.76  122.12  123.29  123.08  123.01  123.49   123.6
  125.52  126.12  126.73
  4596.3  4726.3  4821.2  4871.2  4875.6  4891.2  4931.2  4941.2  4951.2  4965.6
  4971.2 4972.91    4973 5026.89    5027  5034.2  5054.2  5074.2  5094.2  5124.2
  5144.2  5154.2  5164.2  5174.2  5184.2  5191.9  5211.9  5231.9  5239.9  5241.9
  5271.9  5281.9  5291.9  5301.9  5309.9  5311.9    5317  5321.9  5331.9  5341.9
    5347  5351.9  5361.9    5367  5371.9  5411.9    5427  5431.9  5441.9  5442.7
    5507    5527  5547.6
  130.13  126.85   124.9  123.49  123.16  122.24  121.61  121.45   121.3  121.07
  121.07  121.07  121.07  121.05  121.05  121.05  121.05  121.04  121.03  121.03
  121.02  121.02  121.01  121.01     121  120.97  120.91  120.85  120.82  120.84
   121.1  121.21  121.31  121.43  121.57  121.54  121.45  121.57  121.82  122.06
  122.19  122.49  123.09   123.4  123.55  124.75  125.21  125.29  125.48  125.49
  126.79  126.17  126.71
   130.1  126.81  124.86  123.45  123.12  121.95  120.91  121.33  120.28  117.74
  116.75  116.54  119.54  119.52  116.84  117.86  119.02  120.87  120.83  116.98
  117.29  118.67  118.92  118.54  118.72  119.16   119.1  119.49  119.27  119.22
  119.94  119.77  120.27  120.11  120.73  120.88   120.7  120.53  120.99  120.86
  121.18  121.48  121.34  121.71  122.07  123.24  123.03  122.96  123.44  123.55
  125.47  126.07  126.68
Pier Skew, UpSta & Num, DnSta & Num=  ,4990.2, 2 ,4990.2, 2 , 0 , 0 , 0 ,,
       1       1
   112.7  120.58
       1       1
  112.65  120.53
Pier Skew, UpSta & Num, DnSta & Num=  ,5009.7, 2 ,5009.7, 2 , 0 , 0 , 0 ,,
       1       1
   112.7  120.58
       1       1
  112.65  120.53
Abutment Skew #Up #Dn= , 2 , 2
  4972.8  4980.5
  119.59  115.67
  4972.8  4980.5
  119.54  115.62
Abutment Skew #Up #Dn= , 2 , 2
  5019.5 5027.09
  115.26  119.57
  5019.5 5027.09
  115.21  119.52
BR Coef= 1 , 1 , 0 ,1.25, 0 ,,,0.8,0,2,0,
WSPro=,,,, 1 ,,,, 0 ,,,, 0 ,,,,-1 ,-1 ,-1 , 0 , 0 , 0 , 0 , 0
BR U #Sta/Elev= 71
  4596.3  130.15  4609.2  129.82  4639.2  129.06  4689.2   127.8  4699.2  127.55
  4726.3  126.86  4821.2  124.91  4845.6  124.22  4855.6  123.94  4871.2   123.5
  4875.6  123.17  4891.2     122  4931.2  120.96  4941.2  121.38  4951.2  120.33
  4965.6  117.79  4971.2   116.8 4972.91  116.59    4973  116.58  4980.5  115.67
  4981.2  115.59  4981.5     115    4988   113.7    5012   113.7  5018.5     115
  5019.5  115.26  5024.2  116.49 5026.89  116.87    5027  116.89  5034.2  117.91
  5054.2  119.07  5074.2  120.92  5094.2  120.88  5124.2  117.03  5144.2  117.34
  5154.2  118.72  5164.2  118.97  5174.2  118.59  5179.9  118.69  5184.2  118.77
  5191.9  119.21  5211.9  119.15  5231.9  119.54  5239.9  119.32  5241.9  119.27
  5259.9   119.7  5271.9  119.99  5281.9  119.82  5291.9  120.32  5299.9  120.19
  5301.9  120.16  5309.9  120.78  5311.9  120.93    5317  120.75  5321.9  120.58
  5331.9  121.04  5341.9  120.91    5347  121.23  5351.9  121.53  5361.9  121.39
    5367  121.76  5371.9  122.12  5411.9  123.29    5427  123.08  5431.9  123.01
    5437  123.25  5441.9  123.49  5442.7   123.6    5507  125.52    5527  126.12
  5547.6  126.73
BR U #Mann= 3
  4596.3     .14  4981.5    .048  5018.5     .14
BR U Banks=4981.5,5018.5
BR D #Sta/Elev= 71
  4596.3   130.1  4609.2  129.77  4639.2  129.01  4689.2  127.75  4699.2   127.5
  4726.3  126.81  4821.2  124.86  4845.6  124.17  4855.6  123.89  4871.2  123.45
  4875.6  123.12  4891.2  121.95  4931.2  120.91  4941.2  121.33  4951.2  120.28
  4965.6  117.74  4971.2  116.75 4972.91  116.54    4973  116.53  4980.5  115.62
  4981.2  115.54  4981.5  114.95    4988  113.65    5012  113.65  5018.5  114.95
  5019.5  115.21  5024.2  116.44 5026.89  116.82    5027  116.84  5034.2  117.86
  5054.2  119.02  5074.2  120.87  5094.2  120.83  5124.2  116.98  5144.2  117.29
  5154.2  118.67  5164.2  118.92  5174.2  118.54  5179.9  118.64  5184.2  118.72
  5191.9  119.16  5211.9   119.1  5231.9  119.49  5239.9  119.27  5241.9  119.22
  5259.9  119.65  5271.9  119.94  5281.9  119.77  5291.9  120.27  5299.9  120.14
  5301.9  120.11  5309.9  120.73  5311.9  120.88    5317   120.7  5321.9  120.53
  5331.9  120.99  5341.9  120.86    5347  121.18  5351.9  121.48  5361.9  121.34
    5367  121.71  5371.9  122.07  5411.9  123.24    5427  123.03  5431.9  122.96
    5437   123.2  5441.9  123.44  5442.7  123.55    5507  125.47    5527  126.07
  5547.6  126.68
BR D #Mann= 3
  4596.3     .14  4981.5    .048  5018.5     .14
BR D Banks=4981.5,5018.5
BC Design=,, 0 ,, 0 ,,,,,,
BC HTab HWMax=130.09
BC Use User HTab Curves=0
BC User HTab FreeFlow(D)= 0

Type RM Length L Ch R = 1 ,81606.1 ,397.5,397.5,397.5
BEGIN DESCRIPTION:
Downstream Section of Bridge/Culvert/Weir
END DESCRIPTION:
#Sta/Elev= 30
  4596.3  130.08  4821.2  124.84  4871.2  123.43  4891.2  121.93  4931.2  120.89
  4941.2  121.31  4951.2  120.26  4971.2  116.73  4981.2  115.52  4981.5  114.93
    4988  113.63    5012  113.63  5018.5  114.93  5024.2  116.42  5034.2  117.84
  5074.2  120.85  5094.2  120.81  5124.2  116.96  5144.2  117.27  5154.2  118.65
  5164.2   118.9  5174.2  118.52  5191.9  119.14  5241.9   119.2  5301.9  120.09
  5311.9  120.86  5341.9  120.84  5411.9  123.22  5431.9  122.94  5547.6  126.66
#Mann= 3 , 1 , 0
  4596.3     .14       0  4981.5    .048       0  5018.5     .14       0
#XS Ineff= 2 , 0
       0    4963   121.1    5037       0   120.8
Permanent Ineff=
       F       F
Bank Sta=4981.5,5018.5
XS Rating Curve= 0 ,0
Exp/Cntr=0.5,0.3

Type RM Length L Ch R = 1 ,81208.6 ,478.2,478.2,478.2
BEGIN DESCRIPTION:
Black Creek US 158.0
END DESCRIPTION:
#Sta/Elev= 30
    4494  130.07    4544   129.1    4684  122.71    4834  119.28    4854  117.75
    4864  118.05    4914  116.47    4924  116.59    4934  117.29    4944  116.72
    4954  116.94    4964  117.84    4974  117.71  4992.3  115.93  4994.3  112.93
  5005.7  112.93  5007.7  115.93  5030.2  117.27  5050.2  117.64  5060.2  117.47
  5080.2  118.17  5330.2   118.3  5340.2  117.76  5360.2  118.02  5370.2  120.53
  5390.2  123.09  5400.2  123.75  5430.2  122.44  5670.2  126.27  5722.7  128.71
#Mann= 3 , 1 , 0
    4494     .14       0  4992.3    .048       0  5007.7     .14       0
Bank Sta=4992.3,5007.7
XS Rating Curve= 0 ,0
Exp/Cntr=0.3,0.1

Type RM Length L Ch R = 1 ,80730.4 ,769.2,769.2,769.2
BEGIN DESCRIPTION:
Black Creek US 157.0
END DESCRIPTION:
#Sta/Elev= 25
  4406.8  127.98  4646.8  118.64  4886.8   116.2  4936.8  116.19  4976.8  116.88
  4986.8  116.21  4992.3  114.12  4994.3  112.12  5005.7  112.12  5007.7  114.12
  5009.5     114  5029.5  115.51  5109.5  116.94  5139.5   116.7  5169.5  119.72
  5179.5  120.19  5199.5  119.02  5209.5  119.79  5219.5  123.33  5229.5  125.48
  5249.5  125.62  5269.5  125.02  5319.5  127.24  5389.5  127.75  5418.8  128.45
#Mann= 3 , 1 , 0
  4406.8     .14       0  4992.3    .048       0  5007.7     .14       0
Bank Sta=4992.3,5007.7
XS Rating Curve= 0 ,0
Exp/Cntr=0.3,0.1

Type RM Length L Ch R = 1 ,79961.2 ,785.4,785.4,785.4
BEGIN DESCRIPTION:
Black Creek US 156.0
END DESCRIPTION:
#Sta/Elev= 30
  4378.5  123.03  4428.5  121.52  4448.5  121.85  4468.5  120.54  4578.5  120.02
  4638.5  118.61  4688.5  116.71  4748.5  115.62  4758.5  114.84  4798.5  114.15
  4808.5  114.78  4818.5   114.8  4828.5  114.33  4838.5  114.71  4848.5  114.12
  4858.5   114.2  4868.5  114.84  4958.5  115.18  4978.5  114.48  4992.3  113.19
  4994.3  111.19  5005.7  111.19  5007.7  113.19  5053.9  116.24  5193.9  114.08
  5343.9   114.6  5393.9  116.71  5413.9  118.71  5433.9  119.37  5451.9  121.23
#Mann= 3 , 1 , 0
  4378.5     .14       0  4992.3    .048       0  5007.7     .14       0
Bank Sta=4992.3,5007.7
XS Rating Curve= 0 ,0
Exp/Cntr=0.3,0.1

Type RM Length L Ch R = 1 ,79175.8 ,647.8,647.8,647.8
BEGIN DESCRIPTION:
Black Creek US 154.0
END DESCRIPTION:
#Sta/Elev= 30
  3974.8  122.65  3994.8  122.26  4054.8  122.37  4104.8  120.93  4144.8  120.21
  4214.8  119.77  4274.8  118.81  4304.8  119.15  4404.8  117.37  4634.8  115.41
  4714.8   113.3  4764.8  114.11  4854.8  112.66  4874.8  113.31  4884.8  113.04
  4974.8  113.75    4992  112.07    4994  110.07  5006.1  110.07  5008.1  112.07
  5045.5  113.79  5065.5  113.32  5115.5  114.19  5135.5  113.53  5195.5  113.53
  5215.5   114.1  5225.5  115.58  5255.5  122.63  5295.5  124.57    5327  125.04
#Mann= 3 , 1 , 0
  3974.8     .14       0    4992    .048       0  5008.1     .14       0
Bank Sta=4992,5008.1
XS Rating Curve= 0 ,0
Exp/Cntr=0.3,0.1

Type RM Length L Ch R = 1 ,78528.0 ,769,769,769
BEGIN DESCRIPTION:
Black Creek US 153.0
END DESCRIPTION:
#Sta/Elev= 30
  3922.8  122.51  3952.8  122.16  3982.8  120.98  4012.8  120.93  4072.8  119.25
  4092.8  119.43  4172.8  116.49  4202.8  115.99  4332.8  115.05  4342.8  115.52
  4399.9  115.37  4492.8  114.64  4522.8  115.17  4552.8  114.54  4592.8  114.77
  4602.8  114.32  4792.8  113.94  4812.8  113.07  4922.8  112.02  4932.8  112.53
    4992   111.6    4994   109.6    5006   109.6    5008   111.6  5400.3  112.61
  5460.3  111.41  5500.3  112.43  5540.3  118.03  5550.3  119.89  5603.8  124.12
#Mann= 4 , 1 , 0
  3922.8      10       0  4399.9     .14       0    4992    .048       0
    5008     .14       0
Bank Sta=4992,5008
XS Rating Curve= 0 ,0
Exp/Cntr=0.3,0.1

Type RM Length L Ch R = 1 ,77759.0 ,787.5,787.5,787.5
BEGIN DESCRIPTION:
Black Creek US 152.0
END DESCRIPTION:
#Sta/Elev= 30
  4069.1  120.73  4209.1  118.78  4219.1  118.15  4239.1  117.73  4359.1  119.56
  4479.1  116.61  4489.1  116.04  4499.1  116.04  4509.1  115.18  4529.1  115.16
  4549.1  114.19  4579.1  114.83  4599.1  113.75  4609.1  114.54  4669.1  112.79
  4779.1  112.27  4889.1  110.49  4991.6  111.95  4993.6  107.95  5006.3  107.95
  5008.3  111.95  5186.1  112.61  5196.1  111.62  5276.1  111.34  5466.1  112.68
  5476.1  113.19  5496.1  115.85  5516.1  117.91  5566.1  119.83  5595.8  122.13
#Mann= 3 , 1 , 0
  4069.1     .15       0  4991.6    .049       0  5008.3     .15       0
Bank Sta=4991.6,5008.3
XS Rating Curve= 0 ,0
Exp/Cntr=0.3,0.1

Type RM Length L Ch R = 1 ,76971.5 ,578.8,578.8,578.8
BEGIN DESCRIPTION:
Black Creek US 151.0
END DESCRIPTION:
#Sta/Elev= 30
  4084.9  119.38  4164.9     118  4224.9  117.51  4414.9  114.03  4454.9  114.82
  4494.9  112.06  4504.9  110.84  4574.9  111.94  4674.9  109.27  4804.9  109.04
  4894.9  109.58  4904.9  110.47  4954.9  110.51  4991.7  109.42  4993.7  105.42
  5006.4  105.42  5008.4  109.42  5026.6  109.79  5096.6  109.52  5126.6  110.92
  5146.6  109.67  5266.6  110.23  5296.6  111.43  5326.6  110.38  5336.6  110.59
  5356.6  112.01  5416.6  112.02  5446.6  113.69  5466.6  116.52  5485.2  117.01
#Mann= 3 , 1 , 0
  4084.9     .15       0  4991.7    .049       0  5008.4     .15       0
Bank Sta=4991.7,5008.4
XS Rating Curve= 0 ,0
Exp/Cntr=0.3,0.1

Type RM Length L Ch R = 1 ,76392.7 ,671.1,671.1,671.1
BEGIN DESCRIPTION:
Black Creek US 149.0
END DESCRIPTION:
#Sta/Elev= 30
  4021.2  118.51  4201.2  118.36  4411.2  113.38  4471.2  112.76  4491.2  111.16
  4541.2  111.65  4611.2  111.06  4701.2  110.89  4731.2  110.47  4741.2  110.67
  4881.2  108.66  4951.2  109.27  4961.2  108.94  4981.2  109.39  4991.2  108.91
  4991.6  107.78  4993.6  103.78  5006.3  103.78  5008.3  107.78  5010.8  108.26
  5030.8  109.74  5060.8  109.58  5070.8  108.82  5080.8  109.14  5090.8  108.68
  5120.8  109.52  5230.8  111.65  5269.8  111.44  5339.8   112.3  5477.2   117.6
#Mann= 3 , 1 , 0
  4021.2     .15       0  4991.6    .049       0  5008.3     .15       0
Bank Sta=4991.6,5008.3
XS Rating Curve= 0 ,0
Exp/Cntr=0.3,0.1

Type RM Length L Ch R = 1 ,75721.6 ,722.3,722.3,722.3
BEGIN DESCRIPTION:
Black Creek US 147.0
END DESCRIPTION:
#Sta/Elev= 30
  4029.8  116.59  4079.8  117.36  4199.8  115.62  4319.8   112.8  4349.8  112.78
  4359.8  113.57  4439.8  113.62  4479.8   112.2  4539.8  111.44  4599.9  111.59
  4719.8  110.42  4739.8  108.52  4749.8   109.2  4759.8  108.85  4809.8  110.03
  4959.8  107.72  4989.8  108.18  4991.7  106.07  4993.7  102.07  5006.4  102.07
  5008.4  106.07  5027.3  108.79  5037.3  109.01  5077.3  108.09  5137.3  109.42
  5197.3  108.09  5387.3  109.27  5397.3  110.85  5427.3  113.21  5621.6  122.03
#Mann= 4 , 1 , 0
  4029.8      10       0  4599.9     .15       0  4991.7    .049       0
  5008.4     .15       0
Bank Sta=4991.7,5008.4
XS Rating Curve= 0 ,0
Exp/Cntr=0.3,0.1

Type RM Length L Ch R = 1 ,74999.3 ,531.6,531.6,531.6
BEGIN DESCRIPTION:
Black Creek US 146.0
END DESCRIPTION:
#Sta/Elev= 30
  3519.2  116.45  3629.2  114.74  3659.2  113.48  3699.2  115.26  3759.2  113.07
  3819.2  114.52  4029.2  112.31  4049.2  112.97  4079.2     112  4179.2  112.53
  4219.2  111.87  4229.2  110.71  4279.2  112.51  4499.2  110.89  4549.2  109.84
  4649.9  110.13  4779.2   110.3  4899.2  105.96  4969.2   107.3  4979.2  106.68
    4991  104.59    4993  100.59  5006.9  100.59  5008.9  104.59    5056  106.78
    5136  106.76    5156  107.81    5226  113.43    5296  122.67  5332.6   123.9
#Mann= 4 , 1 , 0
  3519.2      10       0  4649.9     .15       0    4991    .049       0
  5008.9     .15       0
Bank Sta=4991,5008.9
XS Rating Curve= 0 ,0
Exp/Cntr=0.3,0.1

Type RM Length L Ch R = 1 ,74467.7 ,717.1,717.1,717.1
BEGIN DESCRIPTION:
Black Creek US 145.0
END DESCRIPTION:
#Sta/Elev= 30
  3626.3  117.27  3676.3  114.98  3766.3  112.67  3946.3  112.62  3986.3  113.57
  4116.3   112.1  4266.3  107.85  4426.3  107.57  4456.3  106.75  4516.3  107.34
  4586.3  106.45  4606.3  106.93  4656.3  105.49  4756.3  106.48  4796.3   106.4
  4806.3  105.47  4826.3  106.76  4876.3   106.8  4936.3   104.8  4966.3  105.93
    4991  103.99    4993   99.99    5007   99.99    5009  103.99    5050  107.23
    5070  106.63    5290  113.75    5320  115.64    5340  117.76  5401.6  119.49
#Mann= 3 , 1 , 0
  3626.3     .15       0    4991    .049       0    5009     .15       0
Bank Sta=4991,5009
XS Rating Curve= 0 ,0
Exp/Cntr=0.3,0.1

Type RM Length L Ch R = 1 ,73750.6 ,464.3,464.3,464.3
BEGIN DESCRIPTION:
Black Creek US 144.0
END DESCRIPTION:
#Sta/Elev= 30
  3924.5  116.71  3974.5  115.53  4164.5  115.73  4184.5  115.01  4254.5  114.88
  4274.5  113.87  4344.5  114.62  4414.5  112.36  4444.5  110.01  4584.5  107.08
  4604.5  105.95  4714.5  105.52  4734.5  104.14  4744.5   104.8  4914.5  104.52
  4954.5  105.67  4984.5  104.69    4991  103.51    4993   99.51    5007   99.51
    5009  103.51  5034.8  105.21  5174.8  105.57  5214.8   106.8  5234.8  108.25
  5244.8  108.31  5314.8  114.72  5344.8  115.89  5364.8  118.99  5379.7  119.73
#Mann= 3 , 1 , 0
  3924.5     .15       0    4991    .049       0    5009     .15       0
Bank Sta=4991,5009
XS Rating Curve= 0 ,0
Exp/Cntr=0.5,0.3

Type RM Length L Ch R = 1 ,73286.3 ,45,45,45
BEGIN DESCRIPTION:
Upstream Section of Bridge/Culvert/Weir
END DESCRIPTION:
#Sta/Elev= 30
  4385.6  114.52  4495.6  112.88  4555.6  111.04  4605.6  109.04  4635.6  107.27
  4705.6   106.3  4725.6  105.25  4755.6  105.39  4805.6   104.1  4875.6  104.58
  4915.6  103.82  4965.6  104.35  4982.5  104.01    4985   99.01    5015   99.01
  5017.5  104.01  5041.3   105.2  5061.3  105.12  5091.3   106.4  5121.3  105.31
  5131.3  104.62  5171.3   104.1  5231.3  105.87  5251.3   107.3  5261.3  108.34
  5281.3  111.87  5301.3  114.47  5321.3  115.58  5331.3  116.47  5401.3  119.59
#Mann= 3 , 1 , 0
  4385.6     .15       0  4982.5    .049       0  5017.5     .15       0
#XS Ineff= 2 , 0
       0    4962     109    5038       0     109
Permanent Ineff=
       F       F
Bank Sta=4982.5,5017.5
XS Rating Curve= 0 ,0
Exp/Cntr=0.5,0.3

Type RM Length L Ch R = 3 ,73263.8 ,,,
BEGIN DESCRIPTION:
Huckleberry Rd-TOR
Structure ID: Huckleberry Rd
Approximate Survey Structure
END DESCRIPTION:
Bridge Culvert--1,0,-1,-1, 0
Deck Dist Width WeirC Skew NumUp NumDn MinLoCord MaxHiCord MaxSubmerge Is_Ogee
10,25,2.6,0, 56, 56, , , 0.95, 0, 1,1,,
  4385.6  4495.6  4555.6    4584  4605.6  4635.6    4694  4705.6  4725.6    4754
  4755.6    4794  4805.6  4875.6  4915.6  4965.6 4972.41  4972.5    4975  4982.5
    4984    4985    5015  5017.5  5020.8  5021.3    5025 5027.39  5027.5  5041.3
  5060.8  5061.3  5091.3  5100.8  5120.8  5121.3  5131.3  5150.8  5160.8  5171.3
  5200.8  5231.3  5251.3  5260.8  5261.3  5280.8  5281.3  5301.3  5321.3  5330.8
  5331.3  5350.8  5360.8  5370.8  5380.8  5401.3
  114.51  112.87  111.03  109.89  109.42  109.27  108.97  108.94   108.9  108.83
  108.86  109.47  109.52  109.79  109.94  110.14  110.16  110.17  110.17   110.2
  110.21  110.21  110.12  110.11   110.1  110.09  110.06  110.03  110.03  109.89
  109.69  109.69  109.48  109.41  108.99  108.99  108.96  108.91  109.21  109.36
  109.77  109.91     110  110.04  110.07  111.77  111.86  114.46  115.57  116.42
  116.46  117.33  117.77  118.22  118.67  119.58
  114.51  112.87  111.03  109.89  109.03  107.26  106.45  106.29  105.24  105.37
  105.38  104.39  104.09  104.57  103.81  104.34   104.2  108.22  108.22  108.25
  108.26  108.26  108.17  108.16  108.15  108.14  108.11  108.08  104.47  105.19
  105.11  105.11  106.39  106.04  105.32   105.3  104.61  104.36  104.23  104.09
  104.96  105.86  107.29  108.28  108.33  111.77  111.86  114.46  115.57  116.42
  116.46  117.33  117.77  118.22  118.67  119.58
  4385.6  4495.6  4555.6    4584  4605.6  4635.6    4694  4705.6  4725.6    4754
  4755.6    4794  4805.6  4875.6  4915.6  4965.6 4972.41  4972.5    4975  4982.5
    4984    4985    5015  5017.5  5020.8  5021.3    5025 5027.39  5027.5  5041.3
  5060.8  5061.3  5091.3  5100.8  5120.8  5121.3  5131.3  5150.8  5160.8  5171.3
  5200.8  5231.3  5251.3  5260.8  5261.3  5280.8  5281.3  5301.3  5321.3  5330.8
  5331.3  5350.8  5360.8  5370.8  5380.8  5401.3
  114.46  112.82  110.98  109.85  109.42  109.27  108.97  108.94   108.9  108.83
  108.86  109.47  109.52  109.79  109.94  110.14  110.16  110.17  110.17   110.2
  110.21  110.21  110.12  110.11   110.1  110.09  110.06  110.03  110.03  109.89
  109.69  109.69  109.48  109.41  108.99  108.99  108.96  108.91  109.21  109.36
  109.77  109.91     110  110.04  110.07  111.73  111.82  114.42  115.53  116.38
  116.42  117.29  117.73  118.18  118.63  119.53
  114.41  112.77  110.93  109.79  108.93  107.16  106.35  106.19  105.14  105.27
  105.28  104.29  103.99  104.47  103.71  104.24   104.1  108.12  108.12  108.15
  108.16  108.16  108.07  108.06  108.05  108.04  108.01  107.98  104.37  105.09
  105.01  105.01  106.29  105.94  105.22   105.2  104.51  104.26  104.13  103.99
  104.86  105.76  107.19  108.18  108.23  111.67  111.76  114.36  115.47  116.32
  116.36  117.23  117.67  118.12  118.57  119.48
Pier Skew, UpSta & Num, DnSta & Num=  ,4987.5, 2 ,4987.5, 2 , 0 , 0 , 0 ,,
       1       1
      98  109.25
       1       1
    97.9  109.15
Pier Skew, UpSta & Num, DnSta & Num=  ,5012.5, 2 ,5012.5, 2 , 0 , 0 , 0 ,,
       1       1
      98  109.18
       1       1
    97.9  109.08
Abutment Skew #Up #Dn= , 2 , 2
  4972.3    4975
  108.22  104.15
  4972.3    4975
  108.12  104.05
Abutment Skew #Up #Dn= , 2 , 2
    5025 5027.59
  104.33  108.08
    5025 5027.59
  104.23  107.98
BR Coef= 1 , 1 , 0 ,1.25, 0 ,,,0.8,0,2,0,
WSPro=,,,, 1 ,,,, 0 ,,,, 0 ,,,,-1 ,-1 ,-1 , 0 , 0 , 0 , 0 , 0
BR U #Sta/Elev= 56
  4385.6  114.51  4495.6  112.87  4555.6  111.03    4584  109.89  4605.6  109.03
  4635.6  107.26    4694  106.45  4705.6  106.29  4725.6  105.24    4754  105.37
  4755.6  105.38    4794  104.39  4805.6  104.09  4875.6  104.57  4915.6  103.81
  4965.6  104.34 4972.41   104.2  4972.5   104.2    4975  104.15  4982.5     104
    4984     101    4985      99    5015      99  5017.5     104  5020.8  104.12
  5021.3  104.14    5025  104.33 5027.39  104.46  5027.5  104.47  5041.3  105.19
  5060.8  105.11  5061.3  105.11  5091.3  106.39  5100.8  106.04  5120.8  105.32
  5121.3   105.3  5131.3  104.61  5150.8  104.36  5160.8  104.23  5171.3  104.09
  5200.8  104.96  5231.3  105.86  5251.3  107.29  5260.8  108.28  5261.3  108.33
  5280.8  111.77  5281.3  111.86  5301.3  114.46  5321.3  115.57  5330.8  116.42
  5331.3  116.46  5350.8  117.33  5360.8  117.77  5370.8  118.22  5380.8  118.67
  5401.3  119.58
BR U #Mann= 3
  4385.6     .15  4982.5    .049  5017.5     .15
BR U Banks=4982.5,5017.5
BR D #Sta/Elev= 56
  4385.6  114.41  4495.6  112.77  4555.6  110.93    4584  109.79  4605.6  108.93
  4635.6  107.16    4694  106.35  4705.6  106.19  4725.6  105.14    4754  105.27
  4755.6  105.28    4794  104.29  4805.6  103.99  4875.6  104.47  4915.6  103.71
  4965.6  104.24 4972.41   104.1  4972.5   104.1    4975  104.05  4982.5   103.9
    4984   100.9    4985    98.9    5015    98.9  5017.5   103.9  5020.8  104.02
  5021.3  104.04    5025  104.23 5027.39  104.36  5027.5  104.37  5041.3  105.09
  5060.8  105.01  5061.3  105.01  5091.3  106.29  5100.8  105.94  5120.8  105.22
  5121.3   105.2  5131.3  104.51  5150.8  104.26  5160.8  104.13  5171.3  103.99
  5200.8  104.86  5231.3  105.76  5251.3  107.19  5260.8  108.18  5261.3  108.23
  5280.8  111.67  5281.3  111.76  5301.3  114.36  5321.3  115.47  5330.8  116.32
  5331.3  116.36  5350.8  117.23  5360.8  117.67  5370.8  118.12  5380.8  118.57
  5401.3  119.48
BR D #Mann= 3
  4385.6     .15  4982.5    .049  5017.5     .15
BR D Banks=4982.5,5017.5
BC Design=,, 0 ,, 0 ,,,,,,
BC HTab HWMax=119.59
BC Use User HTab Curves=0
BC User HTab FreeFlow(D)= 0

Type RM Length L Ch R = 1 ,73241.3 ,508.5,508.5,508.5
BEGIN DESCRIPTION:
Downstream Section of Bridge/Culvert/Weir
END DESCRIPTION:
#Sta/Elev= 30
  4385.6   114.4  4495.6  112.76  4555.6  110.92  4605.6  108.92  4635.6  107.15
  4705.6  106.18  4725.6  105.13  4755.6  105.27  4805.6  103.98  4875.6  104.46
  4915.6   103.7  4965.6  104.23  4982.5  103.89    4985   98.89    5015   98.89
  5017.5  103.89  5041.3  105.08  5061.3     105  5091.3  106.28  5121.3  105.19
  5131.3   104.5  5171.3  103.98  5231.3  105.75  5251.3  107.18  5261.3  108.22
  5281.3  111.75  5301.3  114.35  5321.3  115.46  5331.3  116.35  5401.3  119.47
#Mann= 3 , 1 , 0
  4385.6     .15       0  4982.5    .049       0  5017.5     .15       0
#XS Ineff= 2 , 0
       0    4962   108.4    5038       0   108.4
Permanent Ineff=
       F       F
Bank Sta=4982.5,5017.5
XS Rating Curve= 0 ,0
Exp/Cntr=0.5,0.3

Type RM Length L Ch R = 1 ,72732.8 ,563.6,563.6,563.6
BEGIN DESCRIPTION:
Black Creek US 69.0
END DESCRIPTION:
#Sta/Elev= 30
  3937.7  115.91  3987.7  114.23  4167.7  112.26  4397.7   111.2  4457.7  109.23
  4737.7   108.5  4807.7  104.92  4837.7  104.32  4857.7  105.14  4917.7  104.39
  4977.7  105.27  4987.7  104.73  4990.5  102.44  4992.5   98.44  5007.6   98.44
  5009.6  102.44  5027.4  102.57  5047.4   103.6  5127.4  103.06  5177.4  103.67
  5217.4  103.42  5237.4  102.88  5271.5  105.08  5301.5  104.73  5341.5  102.86
  5411.5  106.03  5421.5   108.1  5431.5  108.64  5461.5  112.93  5490.3  115.67
#Mann= 3 , 1 , 0
  3937.7     .15       0  4990.5    .049       0  5009.6     .15       0
Bank Sta=4990.5,5009.6
XS Rating Curve= 0 ,0
Exp/Cntr=0.3,0.1

Type RM Length L Ch R = 1 ,72169.2 ,530.7,530.7,530.7
BEGIN DESCRIPTION:
Black Creek US 68.0
END DESCRIPTION:
#Sta/Elev= 30
  3864.3  112.54  3874.3  112.11  3884.3  112.64  3994.3  112.49  4014.3  112.17
  4064.3  112.94  4354.3  108.47  4424.3  105.28  4514.3   104.5  4594.3  104.11
  4634.3  102.81  4990.5  102.05  4992.5   98.05  5007.6   98.05  5009.6  102.05
  5077.7   102.5  5097.7  102.97  5117.7   102.4  5247.7  102.01  5267.7  102.41
  5297.7  102.12  5307.7  102.53  5317.7  103.46  5337.7  103.55  5377.7  106.01
  5407.7  109.19  5427.7  112.34  5437.7  115.38  5447.7  117.85  5454.9  118.28
#Mann= 3 , 1 , 0
  3864.3     .15       0  4990.5    .049       0  5009.6     .15       0
Bank Sta=4990.5,5009.6
XS Rating Curve= 0 ,0
Exp/Cntr=0.3,0.1

Type RM Length L Ch R = 1 ,71638.5 ,490.3,490.3,490.3
BEGIN DESCRIPTION:
Black Creek US 67.0
END DESCRIPTION:
#Sta/Elev= 26
    3889  112.62    3909  112.36    3919  111.89    3959  112.96    3989  112.25
    4139  112.01    4279  112.13    4329  111.75    4349  110.25    4369  110.08
    4469  103.87    4609  102.65    4629  103.11    4739  100.29    4779  100.86
    4859  101.17    4869  100.88    4949  101.56  4990.5  100.43  4992.5   96.43
  5007.6   96.43  5009.6  100.43  5258.3  101.67  5328.3  103.45  5448.3  111.18
  5534.2  113.29
#Mann= 3 , 1 , 0
    3889     .15       0  4990.5    .049       0  5009.6     .15       0
Bank Sta=4990.5,5009.6
XS Rating Curve= 0 ,0
Exp/Cntr=0.3,0.1

Type RM Length L Ch R = 1 ,71148.2 ,463.3,463.3,463.3
BEGIN DESCRIPTION:
Black Creek US 66.0
END DESCRIPTION:
#Sta/Elev= 30
  4109.4  111.24  4219.4  110.73  4329.4  109.49  4389.4     111  4429.4  110.62
  4569.4  102.99  4629.4  102.14  4659.4  102.46  4699.4  100.77  4959.4  101.08
  4990.5    99.6  4992.5    95.6  5007.5    95.6  5009.5    99.6  5025.3  100.96
  5175.3  101.12  5205.3   99.84  5255.3  100.42  5265.3     101  5315.3  100.67
  5335.3  101.11  5345.3  101.84  5365.3  101.48  5385.3  102.27  5475.3  103.72
  5495.3  104.89  5545.3  106.08  5575.3  107.59  5615.3  112.62  5628.5  113.37
#Mann= 3 , 1 , 0
  4109.4     .15       0  4990.5    .049       0  5009.5     .15       0
Bank Sta=4990.5,5009.5
XS Rating Curve= 0 ,0
Exp/Cntr=0.3,0.1

Type RM Length L Ch R = 1 ,70684.9 ,437.7,437.7,437.7
BEGIN DESCRIPTION:
Black Creek US 65.0
END DESCRIPTION:
#Sta/Elev= 30
  4227.3  110.88  4557.3  108.44  4617.3  104.17  4667.3  102.19  4717.3  101.93
  4797.3   99.48  4967.3  100.13  4990.4   98.69  4992.4   94.69  5007.5   94.69
  5009.5   98.69    5010   99.77    5020  100.36    5060    99.9    5070   99.25
    5170   99.91    5210   99.28    5280   99.26    5290   99.66    5300  100.49
    5310  100.16    5320  101.32    5330  104.38    5340  106.34    5350  106.89
    5360  108.77    5380  109.38    5400  111.59    5420  113.14  5459.3  114.71
#Mann= 3 , 1 , 0
  4227.3     .15       0  4990.4    .049       0  5009.5     .15       0
Bank Sta=4990.4,5009.5
XS Rating Curve= 0 ,0
Exp/Cntr=0.3,0.1

Type RM Length L Ch R = 1 ,70247.2 ,914.3,914.3,914.3
BEGIN DESCRIPTION:
Black Creek US 64.0
END DESCRIPTION:
#Sta/Elev= 30
  4340.8  111.92  4570.8  109.38  4680.8  102.79  4700.8  102.16  4740.8  102.23
  4780.8  100.01  4820.8  100.93  4850.8   99.95  4880.8   99.74  4890.8  100.32
  4980.8  100.11  4990.4   98.48  4992.4   94.48  5007.5   94.48  5009.5   98.48
  5037.6   99.98  5127.6   99.37  5137.6    99.9  5167.6    99.8  5187.6   98.47
  5237.6   99.86  5267.6   99.85  5277.6   99.24  5363.9   99.79  5383.9  102.97
  5393.9   103.9  5443.9  104.44  5543.9  110.42  5573.9  113.16  5601.8  113.97
#Mann= 3 , 1 , 0
  4340.8     .15       0  4990.4    .049       0  5009.5     .15       0
Bank Sta=4990.4,5009.5
XS Rating Curve= 0 ,0
Exp/Cntr=0.3,0.1

Type RM Length L Ch R = 1 ,69332.9 ,607.3,607.3,607.3
BEGIN DESCRIPTION:
Black Creek US 63.5
END DESCRIPTION:
#Sta/Elev= 30
  3649.8  108.72  3859.8  108.41  4079.8  103.48  4199.8  102.31  4209.8  101.53
  4349.8  101.71  4419.8  100.18  4459.8  100.89  4519.8   99.89  4559.8  100.48
  4609.8   99.18  4629.8   99.92  4819.8    99.4  4879.8     100  4979.8   99.17
  4990.5   98.17  4992.5   94.17  5007.5   94.17  5009.5   98.17  5009.8   98.88
  5030.6   99.74  5300.6   99.93  5310.6  101.93  5410.6  102.51  5450.6  105.83
  5474.9  106.34  5540.6  104.24  5570.6  105.24  5590.6  109.66  5645.4  114.48
#Mann= 4 , 1 , 0
  3649.8     .15       0  4990.5    .049       0  5009.5     .15       0
  5474.9      10       0
Bank Sta=4990.5,5009.5
XS Rating Curve= 0 ,0
Exp/Cntr=0.3,0.1

Type RM Length L Ch R = 1 ,68725.6 ,635.2,635.2,635.2
BEGIN DESCRIPTION:
Black Creek US 63.0
END DESCRIPTION:
#Sta/Elev= 30
  3746.1  108.75  3816.1  109.11  4216.1  105.64  4346.1   101.4  4386.1  101.24
  4406.1  100.16  4556.1  100.49  4566.1   99.77  4646.1   99.53  4676.1  100.24
  4756.1  100.37  4806.1   99.25  4866.1   99.16  4916.1  100.37  4936.1   99.26
  4946.1   97.68  4990.5   97.73  4992.5   93.73  5007.6   93.73  5009.6   97.73
  5086.5   97.74  5096.5   99.42  5556.5  100.03  5666.5  101.94  5746.5  100.56
  5766.5   99.67  5806.5   100.8  5826.5  102.37  5876.5  109.78  5929.3  112.22
#Mann= 3 , 1 , 0
  3746.1     .15       0  4990.5    .049       0  5009.6     .15       0
Bank Sta=4990.5,5009.6
XS Rating Curve= 0 ,0
Exp/Cntr=0.3,0.1

Type RM Length L Ch R = 1 ,68090.4 ,622.7,622.7,622.7
BEGIN DESCRIPTION:
Black Creek US 62.0
END DESCRIPTION:
#Sta/Elev= 30
  3740.7  109.52  3840.7  108.21  3940.7  105.33  4090.7   104.3  4120.7  103.07
  4210.7  102.57  4230.7  103.71  4690.7    99.2  4710.7   100.1  4820.7   99.97
  4830.7   97.43  4840.7   96.92  4860.7      99  4900.7   99.78  4930.7   96.93
  4990.4   96.97  4992.4   92.97  5007.5   92.97  5009.5   96.97  5134.8   96.99
  5154.8   99.56  5194.8    99.9  5224.8   99.07  5244.8   99.85  5364.8    99.3
  5434.8  100.67  5464.8   99.87  5664.8   99.95  5694.8  103.55  5815.8   108.3
#Mann= 3 , 1 , 0
  3740.7     .15       0  4990.4    .049       0  5009.5     .15       0
Bank Sta=4990.4,5009.5
XS Rating Curve= 0 ,0
Exp/Cntr=0.3,0.1

Type RM Length L Ch R = 1 ,67467.7 ,788,788,788
BEGIN DESCRIPTION:
Black Creek US 61.0
END DESCRIPTION:
#Sta/Elev= 30
  4288.9  108.76  4338.9  107.39  4438.9  102.37  4458.9  100.21  4588.9   99.35
  4608.9   98.63  4668.9   99.12  4748.9   98.06  4788.9   98.48  4838.9   97.89
  4888.9   98.35  4908.9   98.08  4928.9   98.55  4938.9   96.56  4990.5   96.74
  4992.5   92.74  5007.6   92.74  5009.6   96.74    5010   96.56    5060   96.57
    5070   97.49    5080   99.16    5090   99.95    5120   99.25    5180   99.76
    5210  101.56    5290  103.31    5320  103.21    5450  106.12  5482.7  106.36
#Mann= 3 , 1 , 0
  4288.9     .15       0  4990.5    .049       0  5009.6     .15       0
Bank Sta=4990.5,5009.6
XS Rating Curve= 0 ,0
Exp/Cntr=0.3,0.1

Type RM Length L Ch R = 1 ,66679.7 ,539,539,539
BEGIN DESCRIPTION:
Black Creek US 60.0
END DESCRIPTION:
#Sta/Elev= 30
  4268.6  110.84  4428.6  108.05  4618.6  107.66  4680.1  106.92  4720.1   104.7
  4730.1  104.74  4750.1  100.77  4760.1    99.9  4780.1   99.74  4810.1  102.37
  4850.1   99.82  4860.1  100.46  4890.1   99.43  4900.1   98.59  4910.1    96.7
  4930.1   97.25  4960.1    96.3  4982.7   96.45  4984.7   92.45  5015.2   92.45
  5017.2   96.45  5127.2    96.4  5167.2   97.82  5187.2   97.12  5247.2   98.38
  5277.2  101.75  5317.2  103.34  5574.9  106.64  6117.2  103.89    6323  106.32
#Mann= 4 , 1 , 0
  4268.6     .15       0  4982.7    .049       0  5017.2     .15       0
  5574.9      10       0
Bank Sta=4982.7,5017.2
XS Rating Curve= 0 ,0
Exp/Cntr=0.3,0.1

Type RM Length L Ch R = 1 ,66140.7 ,470.5,470.5,470.5
BEGIN DESCRIPTION:
Black Creek US 59.0
END DESCRIPTION:
#Sta/Elev= 26
  4210.2  112.09  4220.2  111.73  4290.2  111.44  4330.2  110.77  4340.2  111.14
  4360.2  110.36  4370.2  109.63  4620.2  108.33  4680.2  107.16  4770.2  103.29
  4820.2   99.21  4910.2   97.14  4920.2   96.45  4982.7   96.25  4984.7   92.25
  5015.2   92.25  5017.2   96.25  5062.4   96.25  5102.4  100.46  5362.4  105.56
  5364.9  105.52  5672.4  100.85  5722.4  101.95  5752.4  102.06  5992.4  109.48
  6111.9  110.66
#Mann= 4 , 1 , 0
  4210.2     .15       0  4982.7    .049       0  5017.2     .15       0
  5364.9      10       0
Bank Sta=4982.7,5017.2
XS Rating Curve= 0 ,0
Exp/Cntr=0.5,0.3

Type RM Length L Ch R = 1 ,65670.2 ,44,44,44
BEGIN DESCRIPTION:
Upstream Section of Bridge/Culvert/Weir
END DESCRIPTION:
#Sta/Elev= 30
  4307.1  113.07  4347.1  111.82  4417.1  111.33  4437.1  110.33  4527.1  111.27
  4637.1  109.36  4697.1  104.84  4747.1  103.17  4797.1   98.37  4897.1   97.65
  4937.1   96.11  4971.5   96.21  4972.5   91.91  5027.5   91.91  5028.5   96.21
  5156.3   97.74  5206.3   99.56  5326.3   98.66  5396.3   96.85  5406.3   97.55
  5486.3   97.04  5546.3   97.65  5581.4   96.73  5771.4   96.89  5978.1   100.9
  6078.1  104.83  6138.1   105.4  6168.1  106.98  6358.1  109.56  6382.6  108.75
#Mann= 3 , 1 , 0
  4307.1     .15       0  4971.5    .049       0  5028.5     .15       0
#XS Ineff= 2 , 0
       0    4959     103    5041       0   102.8
Permanent Ineff=
       F       F
Bank Sta=4971.5,5028.5
XS Rating Curve= 0 ,0
Exp/Cntr=0.5,0.3
