--- DTL_Bloomery_Swp_T3.prj (project) ---

Proj Title=DTL_Bloomery_Swp_T3
Current Plan=p01
Default Exp/Contr=0.3,0.1
English Units
Geom File=g01
Flow File=f01
Flow File=f02
Plan File=p01
Plan File=p02
Y Axis Title=Elevation
X Axis Title(PF)=Main Channel Distance
X Axis Title(XS)=Station
BEGIN DESCRIPTION:
END DESCRIPTION:
DSS Export Rating Curves= 0
DSS Export Rating Curve Sorted= 0
DSS Export Volume Flow Curves= 0
DXF OffsetX= 0
DXF OffsetY= 0
DXF ScaleX= 1
DXF ScaleY= 10

--- DTL_Bloomery_Swp_T3.p01 (plan) ---

Plan Title=DTL_Bloomery_Swp_T3
Program Version=4.00
Short Identifier=Multi Profile
Geom File=g01
Flow File=f01
Subcritical Flow
K Sum by GR= 0
Std Step Tol= 0.01
Critical Tol= 0.01
Num of Std Step Trials= 20
Max Error Tol= 0.3
Flow Tol Ratio= 0.001
Split Flow NTrial= 30
Split Flow Tol= 0.02
Split Flow Ratio= 0.02
Log Output Level= 0
Friction Slope Method= 1
Unsteady Friction Slope Method= 2
Unsteady Bridges Friction Slope Method= 1
Parabolic Critical Depth
Global Vel Dist= 0 , 0 , 0
Global Log Level= 0
CheckData=True
Encroach Param=-1 ,10,10, 2
Encroach River=Bloomery Swamp
Encroach Reach=Trib 3
Encroach Node=10437
       1     498     575
Encroach Node=10181
       1     537     613
Encroach Node=9873
       1     428     502
Encroach Node=9459
       1     490     565
Encroach Node=9217
       1     425     505
Encroach Node=8973
       1     731     853
Encroach Node=8787
       1     765     887
Encroach Node=8567
       1     687     795
Encroach Node=8247
       1     300     394
Encroach Node=7767
       1     221     304
Encroach Node=7384
       1     380     451
Encroach Node=6880
       1     318     362
Encroach Node=6523
       1     474     541
Encroach Node=6357
       1  652.25     810
Encroach Node=6286
       1  677.34     835
Encroach Node=6174
       1     642     905
Encroach Node=5798
       1   617.5    1020
Encroach Node=5470
       1     670    1070
Encroach Node=5222
       1     419     463
Encroach Node=4746
       1     330     405
Encroach Node=4336
       1     420     480
Encroach Node=3896
       1     422     476
Encroach Node=3492
       1     303     360
Encroach Node=2983
       1     465     526
Encroach Node=2476
       1     180     250
Encroach Node=2326
       1  251.75     327
Encroach Node=2261
       1  253.24     327
Encroach Node=2084
       1     180     214
Encroach Node=1851
       1     310     346
Encroach Node=1708
       1     869     911
Encroach Node=1477
       1     850  888.25
Encroach Node=1284
       1     675     775
Encroach Node=831
       1     230     335
Encroach Node=578
       1   69.18     215
Encroach Node=233
       1  139.55     280
Encroach Node=58
       1     370     490
Computation Interval=1HOUR
Output Interval=1HOUR
Run HTab= 0
Run UNet= 0
Run PostProcess= 0
Run WQNet= 0
UNET Theta= 1
UNET Theta Warmup= 1
UNET ZTol= 0.02
UNET ZSATol= 0.05
UNET MxIter= 20
UNET MaxInSteps= 0
UNET DtIC= 0
UNET DtMin= 0
UNET MaxCRTS= 20
UNET WFStab= 2
UNET SFStab= 1
UNET WFX= 1
UNET SFX= 1
UNET DSS MLevel= 4
UNET DZMax Abort= 100
UNET Convert EG Bridges= 0
UNET Use Existing IB Tables=-1
UNET Froude Reduction=False
UNET Froude Limit= 1
UNET Froude Power= 10
UNET Time Slicing=0,0, 5
Instantaneous Interval=1HOUR
Write IC File= 0
Echo Input=False
Echo Output=False
Write Detailed= 0
Detailed Automatic Start=False, 10
WQ ULTIMATE=-1
WQ Max Comp Step=1HOUR
WQ Output Interval=15MIN
WQ Output Selected Increments= 0
WQ Output face flow=0
WQ Output face velocity=0
WQ Output face area=0
WQ Output face dispersion=0
WQ Output cell volume=0
WQ Output cell surface area=0
WQ Output cell continuity=0
WQ Output face conc=0
WQ Output face dconc_dx=0
WQ Output face courant=0
WQ Output face peclet=0
WQ Output face adv mass=0
WQ Output face disp mass=0
WQ Output cell mass=0
WQ Output cell source sink temp=0
WQ Output cell source sink nsm=0
WQ Output MaxMinRange=-1
WQ Daily Max Min Mean=-1
WQ Daily Range=0
WQ Daily Time=0
WQ Create Restart=0
WQ Fixed Restart=0
WQ System Summary=False
Sorting and Armoring Iterations= 10
XS Update Threshold= 0.02
Hydraulics Update Threshold= 0.02
Energy Slope Method= 1
Volume Change Method= 0
XS Weighting Method= 0
Number of US Weighted Cross Sections= 1
Number of DS Weighted Cross Sections= 1
Upstream XS Weight=0.25
Main XS Weight=0.5
Downstream XS Weight=0.25
Number of DS XS's Weighted with US Boundary= 1
Upstream Boundary Weight= 1
Weight of XSs Associated with US Boundary= 0
Number of US XS's Weighted with DS Boundary= 1
Downstream Boundary Weight= 0.5
Weight of XSs Associated with DS Boundary= 0.5
Sediment Output Level= 4
Mass or Volume Output= 0
Output Increment Type= 1
Profile and TS Output Increment= 10
XS Output Flag= 0
XS Output Increment= 10
Disregard all LS=0
Disregard all Conn=0
Disregard all Breaches=0
Disregard all Pumps=0

--- DTL_Bloomery_Swp_T3.p02 (plan) ---

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Plan Title=DTL_Bloomery_Swp_T3_Future
Short Identifier=Future
Geom File=g01
Flow File=f02
Encroach Param=-1 ,0,0, 0

--- DTL_Bloomery_Swp_T3.f01 (steady flow) ---

Flow Title=DTL_Bloomery_Swp_T3
Program Version=4.00
Number of Profiles= 6
Profile Names=100-yr,FW,10-yr,25-yr,50-yr,500-yr
River Rch & RM=Bloomery Swamp,Trib 3          ,10437
     680     680     280     420     540    1100
River Rch & RM=Bloomery Swamp,Trib 3          ,3492
     750     750     310     460     600    1210
Boundary for River Rch & Prof#=Bloomery Swamp,Trib 3          , 1
Up Type= 0
Dn Type= 3
Dn Slope=3.714286E-03
Boundary for River Rch & Prof#=Bloomery Swamp,Trib 3          , 2
Up Type= 0
Dn Type= 3
Dn Slope=3.714286E-03
Boundary for River Rch & Prof#=Bloomery Swamp,Trib 3          , 3
Up Type= 0
Dn Type= 3
Dn Slope=3.714286E-03
Boundary for River Rch & Prof#=Bloomery Swamp,Trib 3          , 4
Up Type= 0
Dn Type= 3
Dn Slope=3.714286E-03
Boundary for River Rch & Prof#=Bloomery Swamp,Trib 3          , 5
Up Type= 0
Dn Type= 3
Dn Slope=3.714286E-03
Boundary for River Rch & Prof#=Bloomery Swamp,Trib 3          , 6
Up Type= 0
Dn Type= 3
Dn Slope=3.714286E-03
DSS Import GetInterval= 0
DSS Import GetPeak= 0
DSS Import FillOption= 0

--- DTL_Bloomery_Swp_T3.f02 (steady flow) ---

Flow Title=DTL_Bloomery_Swp_T3_Future
Program Version=4.00
Number of Profiles= 3
Profile Names=100-yr-10%,100-yr-20%,100-yr-35%
River Rch & RM=Bloomery Swamp,Trib 3          ,10437
    1190    1520    1860
River Rch & RM=Bloomery Swamp,Trib 3          ,3492
    1310    1680    2050
Boundary for River Rch & Prof#=Bloomery Swamp,Trib 3          , 1
Up Type= 0
Dn Type= 3
Dn Slope=3.714286E-03
Boundary for River Rch & Prof#=Bloomery Swamp,Trib 3          , 2
Up Type= 0
Dn Type= 3
Dn Slope=3.714286E-03
Boundary for River Rch & Prof#=Bloomery Swamp,Trib 3          , 3
Up Type= 0
Dn Type= 3
Dn Slope=3.714286E-03
DSS Import GetInterval= 0
DSS Import GetPeak= 0
DSS Import FillOption= 0

--- DTL_Bloomery_Swp_T3.g01 (geometry) ---

Geom Title=DTL_Bloomery_Swp_T3
Program Version=4.00

River Reach=Bloomery Swamp  ,Trib 3
Reach XY= 30
 2301129.8178698  741050.8927999 2301188.2432718  740791.1456386
 2301342.9638176  740762.0284879 2301550.2094194  740532.5168297
 2301877.9200956  739999.2733253 2301896.1896803  739496.8597451
 2301991.5340756  739442.0509909 2302032.0697168  739315.3057469
 2301900.7570765   738696.423564 2301952.1402835  738462.3445096
 2301795.1360398  738286.4997566 2301838.5263035  738210.5667951
 2301797.4197378  738108.3713054 2301663.8233995  738050.1370041
 2301634.7062488  737897.7001565 2301522.0834837  737798.3661559
 2301427.4606469  737180.0480312 2301240.2946135  737070.1628534
 2301228.2079885  736217.4692855  2300979.855821  735865.2088549
 2300707.5248236  735725.3323468 2299954.4753779  734966.5736559
 2299634.1867205  734535.5256411  2299518.274238  733914.9536568
 2299423.5155716  733735.6603845 2299477.1824767  733519.2799903
 2299622.7682301  733406.8078593 2299646.1761355  733162.4521635
 2299488.6009672  732884.9828454  2299270.755986  732816.1924755

Type RM Length L Ch R = 1 ,10437   ,218.04,255.86,254.33
XS GIS Cut Line= 3
 2301622.7233446  741249.9842852 2300967.5829108  740958.5584768
 2300573.1469479  740696.7957844
#Sta/Elev= 30
       0  154.02   81.91  154.21  118.85  153.64  149.79  154.13  172.74  152.96
     211  153.35  271.48  151.88  317.77  152.53  397.27   152.1  464.53  149.45
  497.36  146.63  512.98  146.13  528.72  145.27  546.08  146.12  635.28  147.98
  640.41  147.42  684.53  149.48  712.71  149.49  744.44  150.78  755.39  150.61
  789.98  152.44  816.21  151.77  836.98  152.54  895.53  153.12 1037.83  153.16
 1070.83  153.61 1089.72  155.08 1102.86   156.1 1121.96   155.1 1190.43  155.99
#Mann= 5 ,-1 , 0
       0     .09       0  512.98     .05       0  546.08     .09       0
  712.71      .1       0 1089.72     .09       0
Bank Sta=512.98,546.08
XS Rating Curve= 0 ,0
Exp/Cntr=0.3,0.1

Type RM Length L Ch R = 1 ,10181   ,245.16,308.83,245.49
XS GIS Cut Line= 3
 2301689.1289149  741099.1169841 2301320.6877448  740878.8320517
 2300778.7478226  740520.1380025
#Sta/Elev= 30
       0  154.14   17.73  153.91   26.84  154.54   43.22  153.35   84.76  154.11
   91.32     153  106.18  152.67  130.03  153.53  244.34  152.93   311.9  151.02
  335.81   151.4  369.54  150.82  389.05  149.48   427.3   148.8  486.89  146.29
  529.09   146.1  539.68  147.47  555.91  147.63  570.72  147.36  582.01  146.15
  589.03  145.07  598.29  146.03  645.88  151.71  695.63  152.78  740.08   152.5
  761.67  153.16  783.39  152.81  824.05  153.73  853.12  153.37 1079.16  155.53
#Mann= 5 ,-1 , 0
       0     .09       0  582.01     .05       0  598.29     .09       0
  695.63      .1       0  761.67    .045       0
Bank Sta=582.01,598.29
XS Rating Curve= 0 ,0
Exp/Cntr=0.3,0.1

Type RM Length L Ch R = 1 ,9873    ,414.06,413.64,410.81
XS GIS Cut Line= 3
 2301810.4123002  740894.3631061 2301237.4670672  740548.6202931
 2300970.7511829  740370.8097035
#Sta/Elev= 30
       0  153.55   37.49  154.06   44.47  153.22    67.2  153.62  114.71  153.08
  160.08  152.13  167.35  152.73  296.72  151.13  345.78   149.5  371.83  147.15
  379.21  147.31  384.55  146.46   397.3  146.34  415.59  144.97   439.2  144.96
   453.8  145.67  458.37  145.24  464.55  144.42  474.92  145.15  515.59  145.87
   578.6  148.37  585.24  148.08  627.21  149.97  651.15  150.36  663.68  151.06
  685.65  150.58  777.24  152.78  806.54  152.56  881.66  154.33  989.73  155.79
#Mann= 6 ,-1 , 0
       0     .09       0    67.2     .04       0  114.71     .09       0
  458.37     .05       0  474.92     .09       0  651.15    .045       0
#XS Ineff= 2 , 0
       0                     595       0
Permanent Ineff=
       F       F
Bank Sta=458.37,474.92
XS Rating Curve= 0 ,0
Exp/Cntr=0.3,0.1

Type RM Length L Ch R = 1 ,9459    ,239.14,241.96,244.67
XS GIS Cut Line= 4
 2302147.2435973  740529.8851233 2301874.3242121  740444.1104594
 2301566.3151916  740286.2071008 2301168.6326587  740212.1289819
#Sta/Elev= 30
       0  153.31   12.48  152.99   27.35  153.59   39.46  152.97  124.67  152.59
   304.8  147.75  359.37  146.68  405.94  146.52  421.64  145.53  488.24  144.45
   513.6  145.39   530.7  144.69  549.13  143.96  554.26  144.67  583.15   147.3
  600.21  149.61  615.09  149.86  639.21  151.11  691.37  151.38  715.97   151.8
   731.8  153.05  744.58152.7372  766.56  153.82  817.04  154.82   824.2  154.49
  862.53  153.62   888.3  155.22   957.8  156.24  966.35   155.9 1036.73  157.27
#Mann= 7 ,-1 , 0
       0     .04       0  421.64     .08       0   530.7     .05       0
  554.26     .09       0  615.09    .045       0  744.58     .09       0
   824.2    .045       0
#XS Ineff= 2 , 0
       0     350                       0
Permanent Ineff=
       F       F
Bank Sta=530.7,554.26
XS Rating Curve= 0 ,0
Exp/Cntr=0.3,0.1

Type RM Length L Ch R = 1 ,9217    ,245.69,243.75,221.93
XS GIS Cut Line= 2
 2302203.0773521  740336.2354222 2301216.1480147  739857.2238691
#Sta/Elev= 30
       0  153.17   39.64  153.17   108.3  152.12  159.73  153.12  173.66  153.21
  189.28  152.26  217.43  152.16  277.18  149.63  295.72  148.36  325.54  147.47
  359.99   145.6  379.75   143.9   388.5  144.59   414.3  143.81  448.14  143.62
     471   143.2  478.96143.6518  509.45  143.33  547.96  143.77  593.33  146.21
   734.5  147.24  743.98   146.7  752.55  147.18  805.01  146.89   828.7   147.3
  853.61  148.64  938.58  149.55  969.89  151.05 1050.71  154.39 1097.03  155.28
#Mann= 5 ,-1 , 0
       0     .04       0  159.73     .08       0  448.14     .05       0
  478.96     .09       0  969.89    .045       0
#XS Ineff= 2 , 0
       0                     655       0
Permanent Ineff=
       F       F
Bank Sta=448.14,478.96
XS Rating Curve= 0 ,0
Exp/Cntr=0.5,0.3

Type RM Length L Ch R = 1 ,8973    ,191.68,185.8,148.53
BEGIN DESCRIPTION:
Surveyed Section
END DESCRIPTION:
XS GIS Cut Line= 6
 2302622.9079108  740264.6172681    2301926.4127     739931.8181
    2301883.2372     739925.9248    2301863.1907     739918.9922
    2301821.6179     739911.8708 2301259.6933909  739624.9930641
#Sta/Elev= 30
       0  153.48  370.16  150.84  437.72  148.58   458.8  149.48  565.89  147.59
  596.79  150.54  603.89  149.06   610.7  150.84  618.13  150.83  677.34  145.54
  686.29  144.69  698.72  146.21  717.97  144.35  757.99  144.84 815.369   143.4
  818.56  142.19 821.751  141.08  830.41   142.2  885.23  143.59 1050.73  143.87
  1149.7  147.61 1167.05  146.09 1196.44  146.73 1272.38  150.17 1326.59  150.89
 1380.35  153.98 1397.87   152.2  1439.1  151.57 1458.23  153.26 1510.24  153.54
#Mann= 9 ,-1 , 0
       0     .04       0  370.16    .035       0  565.89     .08       0
  677.34    .035       0  717.97     .08       0  818.56     .05       0
  830.41     .09       0 1397.87    .045       0  1439.1     .09       0
#XS Ineff= 2 , 0
       0   809.5  148.77   834.5       0  148.77
Permanent Ineff=
       F       F
Bank Sta=818.56,830.41
XS Rating Curve= 0 ,0
Exp/Cntr=0.5,0.3

Type RM Length L Ch R = 2 ,8874    ,,,
BEGIN DESCRIPTION:
Packhouse Road
END DESCRIPTION:
Bridge Culvert--1,0,-1,-1, 0
Deck Dist Width WeirC Skew NumUp NumDn MinLoCord MaxHiCord MaxSubmerge Is_Ogee
87.25,21.5,2.6,0, 17, 17, , , 0.98, 0, 1,1,,
       0    5.49   69.86  194.02  338.25  500.62 762.397 812.876 861.787 909.739
 1149.63 1227.82 1356.25 1411.38 1476.51 1498.48 1510.24
  154.03  154.03  153.83  152.82  151.46  149.68  148.78  148.77  148.94  149.12
  149.82  151.47  153.52  154.21  154.71  154.55  154.55
                                                                                
                                                        
       0    5.49   69.86  194.02  338.25  500.62 762.397 812.876 861.787 909.739
 1149.63 1227.82 1356.25 1411.38 1476.51 1498.48 1510.24
  154.03  154.03  153.83  152.82  151.46  149.68  148.78  148.77  148.94  149.12
  149.82  151.47  153.52  154.21  154.71  154.55  154.55
                                                                                
                                                        
BR Coef=-1 , 0 , 0 ,, 0 ,,,0.8,-1,,0,
WSPro=,,,, 1 ,,,, 0 ,,,, 0 ,,,,-1 ,-1 ,-1 , 0 , 0 , 0 , 0 , 0
Culvert=2,5,8,37.5,0.013,0.4,1,8,1,140.95,822,140.85,857,Culvert #1  , 0 ,79.18
Culvert Bottom n=0.013
BC Design=,, 0 ,, 0 ,,,,,,
BC Use User HTab Curves=0
BC User HTab FreeFlow(D)= 0

Type RM Length L Ch R = 1 ,8787    ,208.03,220.2,227.07
BEGIN DESCRIPTION:
Surveyed Section
END DESCRIPTION:
XS GIS Cut Line= 6
 2302659.9517836  740084.3370871     2301931.569     739725.5434
    2301879.5301     739742.3794    2301871.4575     739742.9916
    2301850.1117     739759.4585 2301296.7372637  739481.7567558
#Sta/Elev= 30
       0  154.32   29.52  152.91   67.53  154.22  142.69  153.58  159.86  155.82
  179.39  152.52  192.29  152.63  319.55  151.65  401.16  149.95  564.16  146.04
  662.71  146.59  756.84  143.27  781.19  143.64 847.525  142.69  850.59   142.1
  856.28  140.86 866.921  142.11 875.015  144.78 901.969  143.32  929.29  144.98
 1056.36  145.49 1094.85  148.37 1144.95   148.1  1166.5  150.21 1212.92  152.12
 1236.77  153.03 1268.44  152.94  1298.6  154.71 1335.68  155.18 1521.28   155.6
#Mann= 7 ,-1 , 0
       0    .065       0  192.29    .045       0  401.16     .09       0
  756.84     .07       0  850.59     .05       0 866.921    .085       0
 1212.92    .045       0
#XS Ineff= 3 ,-1
       0   138.8  164.15   138.8   844.5   144.5   869.5    1600   144.5
Permanent Ineff=
       F       F       F
#Block Obstruct= 1 ,-1
   88.48   138.8 164.149
Bank Sta=850.59,866.921
XS Rating Curve= 0 ,0
Exp/Cntr=0.5,0.3

Type RM Length L Ch R = 1 ,8567    ,281.5,320.35,239.64
XS GIS Cut Line= 2
 2302617.0548249  739730.6212094 2301683.2806424  739459.6512483
#Sta/Elev= 30
       0  154.04    8.43  153.53   43.13  153.62   51.46  153.29  140.77  152.43
  262.93  150.27  300.55  149.97  308.25  149.47  347.98  149.17  418.35  147.53
  440.89  146.29  460.21  145.89  487.83  144.54  564.71  143.26  571.23  143.14
  587.18  141.99  608.13  141.63  637.99   141.3  728.82  141.85  750.61  141.06
   754.9  140.28  764.13  141.03  780.28  142.03  808.36  142.79  820.17  143.61
  843.19  144.31  867.89  146.04  904.56  148.03  913.41  148.08   972.3  152.47
#Mann= 5 ,-1 , 0
       0    .045       0  347.98     .09       0  564.71     .07       0
  750.61     .05       0  764.13    .085       0
#XS Ineff= 2 ,-1
       0   14.34  164.04   14.34     476     146
Permanent Ineff=
       F       F
#Block Obstruct= 1 ,-1
       0   14.34 164.044
Bank Sta=750.61,764.13
XS Rating Curve= 0 ,0
Exp/Cntr=0.3,0.1

Type RM Length L Ch R = 1 ,8247    ,422.63,480.14,384.01
XS GIS Cut Line= 3
 2302388.2967163  739311.3549408 2301884.5000459   739274.311068
 2301652.3584428  739252.0847443
#Sta/Elev= 30
       0   152.2   13.48  151.56   37.53  151.33    42.6   151.1  123.16  149.57
  139.85  149.23  164.06  149.16  204.53  147.16  214.26  146.53  260.99  142.73
  294.11  140.35  323.18  140.62  347.18  139.96  357.15  139.67  367.19  139.93
  389.62  140.43  411.19  141.26  422.34  141.32  441.28  142.67  452.84  143.25
   499.3  144.83  518.85  146.12  553.05  147.89  600.95  148.62  613.29  149.49
  618.52  149.62  641.08  149.61  658.84  150.15  666.38  149.92  738.36  151.95
#Mann= 6 ,-1 , 0
       0    .045       0  123.16    .085       0  204.53     .07       0
  347.18     .05       0  367.19    .085       0  618.52    .045       0
Bank Sta=347.18,367.19
XS Rating Curve= 0 ,0
Exp/Cntr=0.3,0.1

Type RM Length L Ch R = 1 ,7767    ,345.58,382.48,358.86
XS GIS Cut Line= 2
 2302215.4734437  738849.4814798 2301628.6967654  738929.4078712
#Sta/Elev= 30
       0  152.52   39.18  151.39   75.78  150.95  109.41  150.28  141.63  148.54
  167.31  146.62  184.76  143.95  220.06  139.84  228.75  139.61  239.33  139.81
  250.43  139.38  263.72  138.91  274.72  139.38  292.09  140.01  323.03   139.8
  337.63  141.73  343.01  142.12  346.24  142.34  379.35  143.15  422.96  146.78
   447.8  146.44  469.43  147.19  478.74  147.45  486.18   146.4  501.28  146.37
  529.07  148.75  535.45  148.81  550.82  148.67  555.51  148.42   592.2  149.36
#Mann= 5 ,-1 , 0
       0    .085       0  184.76     .07       0  250.43     .05       0
  274.72    .085       0  469.43    .045       0
Bank Sta=250.43,274.72
XS Rating Curve= 0 ,0
Exp/Cntr=0.3,0.1

Type RM Length L Ch R = 1 ,7384    ,382.74,504.48,324.86
XS GIS Cut Line= 2
 2302338.9048858  738528.4944285 2301593.0882463  738545.7815692
#Sta/Elev= 30
       0  152.15   22.12   151.6   56.86  152.12   78.48  151.61  166.15  149.48
  179.11   148.6  195.65  148.22  237.36  146.35  275.14  145.71  301.43  144.17
  322.32  142.22  348.17  141.37  382.29   139.4   403.6  139.03  424.03  138.74
   435.3  139.05  465.28  139.72  489.94  139.73  515.98  141.27  535.02  143.09
  567.12  144.32  590.34  146.08  621.35  149.35   641.4  150.35  650.68150.5354
  686.45  151.83  721.51  152.41  724.52  152.67  736.91  152.85  746.02  152.29
#Mann= 7 ,-1 , 0
       0     .09       0   78.48    .045       0  348.17    .085       0
   403.6     .05       0   435.3    .085       0  567.12    .045       0
  650.68    .085       0
#XS Ineff= 2 , 0
       0     345                       0
Permanent Ineff=
       F       F
Bank Sta=403.6,435.3
XS Rating Curve= 0 ,0
Exp/Cntr=0.3,0.1

Type RM Length L Ch R = 1 ,6880    ,315.42,357.16,291.03
XS GIS Cut Line= 2
 2302143.8071556  738049.3936734 2301560.9835566  738318.5791492
#Sta/Elev= 30
       0  153.31   84.09   152.5  130.55   151.4  144.39  150.45   183.7  148.66
  201.45  147.44  228.04  144.83  271.06  141.79   281.9  140.51  304.75  138.85
  314.55  138.27  332.29  138.65  340.89   137.1   342.5  137.28  347.27  138.64
  361.27  138.21  372.93  138.43  392.91  138.16  423.26  139.02  437.05  140.31
  460.21  141.25   470.7  141.94  480.97  142.15  514.02  144.07  532.81  144.35
  558.18  146.23  570.86  147.68  585.08  148.88  603.84   149.8  641.98  150.88
#Mann= 4 ,-1 , 0
       0    .045       0  332.29     .05       0  347.27    .085       0
  423.26    .045       0
Bank Sta=332.29,347.27
XS Rating Curve= 0 ,0
Exp/Cntr=0.3,0.1

Type RM Length L Ch R = 1 ,6523    ,119.08,165.18,239.46
XS GIS Cut Line= 4
 2302141.3375641  737841.9479855 2301805.4731172  737846.8871686
 2301499.2437685  738039.5153073 2301370.8250094  738185.2212071
#Sta/Elev= 30
       0  151.58    25.5  150.95   62.88   149.4  135.58  149.45  175.51  148.63
  221.25  148.95  233.28  148.73  279.98  149.52  301.93  149.39  319.82  148.64
   335.9  148.47  379.49  145.02  401.37   143.8  413.58  143.57  423.27   142.9
  453.58  142.31  466.16  140.63  473.87  140.45  484.43  136.62  489.51  136.14
  506.38  135.73  530.32  136.61  543.79  139.04  551.12  139.26  572.15  138.36
  578.22   138.5  615.63  139.33  637.44  141.48  712.99   145.4   891.9  149.12
#Mann= 6 ,-1 , 0
       0    .045       0  484.43     .05       0  530.32    .032       0
  543.79    .045       0  578.22    .085       0  637.44    .045       0
Bank Sta=484.43,530.32
XS Rating Curve= 0 ,0
Exp/Cntr=0.5,0.3

Type RM Length L Ch R = 1 ,6357    ,71.85,70.99,56.51
XS GIS Cut Line= 4
 2302230.2428588  737814.7824788 2301538.5265846  737815.5366768
  2301171.269864  737818.2749112 2301082.3371856  737843.7308663
#Sta/Elev= 30
       0  152.87   14.51  152.75    87.9  150.71  151.39  150.27  221.85  150.85
  325.25   150.2  398.29   150.5  536.24  143.62  601.93  141.58  636.73  141.57
  653.28  136.35  655.31  136.26  663.14  136.23  679.22  135.14  691.72  135.26
  694.12  136.13  705.82  136.11  713.93  137.79  719.33     138  736.16  137.52
  769.98  139.05  782.35  138.53  810.46  139.22  825.65  140.29  892.07  141.43
  904.19  141.04  993.29  143.02 1027.09  143.22 1058.98  144.56 1151.49   150.5
#Mann= 4 ,-1 , 0
       0     .09       0   14.51    .045       0  655.31    .032       0
  719.33    .045       0
#XS Ineff= 4 ,-1
       0  652.25     150  652.25  660.75  143.15  697.25  965.98  142.28
  965.98    1200     150
Permanent Ineff=
       F       F       F       F
Bank Sta=663.14,694.12
XS Rating Curve= 0 ,0
Exp/Cntr=0.5,0.3

Type RM Length L Ch R = 2 ,6312    ,,,
BEGIN DESCRIPTION:
Private Drive
END DESCRIPTION:
Bridge Culvert--1,0,-1,-1, 0
Deck Dist Width WeirC Skew NumUp NumDn MinLoCord MaxHiCord MaxSubmerge Is_Ogee
40.25,9.5,2.6,0, 30, 30, , , 0.98, 0, 0.63,0.63,,
       0    6.12   73.15  158.06  175.49  212.95  252.06  330.23  419.24  526.56
  609.07 653.201  663.25  663.25  694.75  694.75 702.698 732.412  781.31  862.76
  929.79 1043.96 1067.96 1110.36 1125.24 1146.74 1147.04 1157.24 1162.34 1167.25
  153.39  153.38  152.19  151.95  151.49  151.36  152.27  150.82  148.92  145.56
  144.08  143.25  143.13  144.13 143.755 142.755  142.66  142.52  142.28  142.31
  142.57  144.76  145.47  148.07  148.88     150  150.02  150.96  151.05  151.33
                                                                                
                                                                                
                                                                                
       0    6.12   73.15  158.06  175.49  212.95  252.06  330.23  419.24  526.56
  609.07 653.201  696.25  696.25 702.698  727.75  727.75 732.412  781.31  862.76
  929.79 1043.96 1067.96 1110.36 1125.24 1146.74 1147.04 1157.24 1162.34 1167.25
  153.39  153.38  152.19  151.95  151.49  151.36  152.27  150.82  148.92  145.56
  144.08  143.25142.7369143.7369  143.66 143.542 142.542  142.52  142.28  142.31
  142.57  144.76  145.47  148.07  148.88     150  150.02  150.96  151.05  151.33
                                                                                
                                                                                
                                                                                
BR Coef=-1 , 0 , 0 ,, 0 ,,,0.8,-1,,0,
WSPro=,,,, 1 ,,,, 0 ,,,, 0 ,,,,-1 ,-1 ,-1 , 0 , 0 , 0 , 0 , 0
Multiple Barrel Culv=1,2,,19,0.024,0.5,1,2,1,138.47,138.18, 4,Culvert #2  , 0 ,35.67
  671.75  704.75     674     707     684     717  686.25  719.25
Culvert Bottom n=0.024
Culvert=1,6,,19,0.012,0.2,1,55,1,135.01,679,134.2,712,Culvert #1  , 0 ,35.67
Culvert Bottom n=0.012
BC Design=,, 0 ,, 0 ,,,,,,
BC Use User HTab Curves=0
BC User HTab FreeFlow(D)= 0

Type RM Length L Ch R = 1 ,6286    ,102.62,112.84,155.42
BEGIN DESCRIPTION:
Surveyed Section
END DESCRIPTION:
XS GIS Cut Line= 6
 2302220.3644927  737760.4514653    2301584.2603     737754.5375
    2301519.8596     737759.1432    2301448.2003     737774.1803
 2301168.6712237   737772.821546 2301060.4291877  737804.4253406
#Sta/Elev= 30
       0  152.84   54.03   153.2   73.71  152.13  128.08  151.82  152.76  150.35
  170.25  150.83  197.91  149.35  264.92  150.96  343.33  149.28  378.06  150.01
  395.83  149.17  416.25  146.94  431.24  146.58  446.33  147.49  472.06  145.09
  498.75  145.12  626.89  141.07 675.327  140.35 699.008  139.76 701.044  138.15
 703.833  134.58 709.608  134.59 723.842  138.13 729.023  140.47 776.567  141.11
  832.62   139.9   847.4  140.98 1031.85   144.6 1052.35  144.08 1168.58  151.91
#Mann= 6 ,-1 , 0
       0    .075       0  498.75    .045       0 675.327    .032       0
 701.044     .05       0 723.842    .032       0 729.023    .045       0
#XS Ineff= 4 ,-1
       0  677.34     150  677.34  693.75  140.18  730.25  950.23  140.18
  950.23    1200     150
Permanent Ineff=
       F       F       F       F
Bank Sta=701.044,723.842
XS Rating Curve= 0 ,0
Exp/Cntr=0.5,0.3

Type RM Length L Ch R = 1 ,6174    ,415.01,375.4,312.03
XS GIS Cut Line= 4
 2302212.9557182  737644.3806638 2301451.1540129  737653.9533218
 2301180.7424221  737657.5308899 2301074.4740268  737674.0157621
#Sta/Elev= 30
       0  150.85   12.85  152.16   38.36  152.65   63.77  151.28   72.12  151.53
  124.24  148.35  139.44  145.57  162.65  144.38  363.44  144.43  394.31  145.02
  412.07  146.27  441.82  145.93  460.04  144.78  493.57  143.83  510.09  144.98
  529.22  144.63  593.09   141.1  618.49  140.81  642.57  138.88  654.02  135.94
  671.77  134.76  726.38  133.75  833.91  134.61  891.56  135.94  900.36  137.21
  904.63  139.05 1067.08  145.03 1093.74  147.18 1120.79  150.72 1139.84  151.62
#Mann= 5 ,-1 , 0
       0    .075       0  460.04    .045       0  642.57    .032       0
  904.63    .032       0  904.63    .045       0
#XS Ineff= 2 , 0
       0     642             905       0
Permanent Ineff=
       F       F
Bank Sta=642.57,904.63
XS Rating Curve= 0 ,0
Exp/Cntr=0.3,0.1

Type RM Length L Ch R = 1 ,5798    ,239.53,328.4,293.19
XS GIS Cut Line= 4
 2302162.8389908  737161.2801395 2301590.6186548  737236.8980628
 2301072.0044353  737399.8911032 2300933.7073101  737548.0665945
#Sta/Elev= 30
       0  154.05   25.48  155.03   39.16  154.24    49.8  152.91   79.27  145.51
   136.7  144.73  180.16  141.87  207.48  143.43  227.46  142.64  238.37   143.7
  251.89  143.79  286.19  142.15  297.53  142.52  366.99  140.88  403.94  141.48
   426.5  140.91  448.27  141.92  509.78  142.67   590.2  140.68  605.67     143
   617.9  141.65  622.31   135.7  695.69  133.35  730.36  133.18  972.26  135.48
 1012.77  136.48 1019.92  138.99 1156.92  142.91 1223.34  147.02 1323.51  149.26
#Mann= 5 ,-1 , 0
       0    .075       0  448.27    .045       0   617.9    .032       0
 1019.92    .032       0 1019.92    .045       0
#XS Ineff= 4 ,-1
       0     519     144     519  605.67     143  605.67   617.5     155
    1020    1400     155
Permanent Ineff=
       F       F       F       F
Bank Sta=617.9,1019.92
XS Rating Curve= 0 ,0
Exp/Cntr=0.5,0.3

Type RM Length L Ch R = 1 ,5470    ,251.27,247.67,240.83
XS GIS Cut Line= 3
 2302146.8608206  737017.8085184   2301486.99526   737029.304434
 2300884.3154797  737123.2968528
#Sta/Elev= 30
       0  154.65   30.01  153.96   82.44  147.39  104.65  146.95  124.08  145.22
  169.47     145  178.26  146.65  188.76   147.1  219.54  144.77  228.81  145.37
  293.99  143.55  434.85  143.18  471.77  142.57  484.73  141.32  502.84  142.17
  528.61  141.21  639.66  141.33  678.92  142.42  714.64  139.97   715.7  137.11
  718.89  135.61  740.51  134.72  912.19  133.21 1001.89  133.89  1049.4   135.5
 1061.77  140.87 1083.51  142.31 1145.99  149.17 1187.95  150.74 1269.93  151.63
#Mann= 7 ,-1 , 0
       0    .075       0  639.66    .045       0  714.64    .032       0
 1061.77    .032       0 1061.77    .045       0 1083.51     .08       0
 1145.99    .045       0
#XS Ineff= 2 , 0
       0  662.78  143.04    1070       0
Permanent Ineff=
       F       F
Bank Sta=714.64,1061.77
XS Rating Curve= 0 ,0
Exp/Cntr=0.5,0.3

Type RM Length L Ch R = 5 ,5434    ,,,
BEGIN DESCRIPTION:
Private Dam w/spillway
END DESCRIPTION:
IW Pilot Flow=0
#Inline Weir SE= 30
       0  154.67   37.44  154.15   62.77  150.76   76.49  147.74  119.04   146.4
  155.54  145.84   176.8  146.96  194.24  147.26  222.73  145.89   300.7  144.47
  389.11  143.75  550.36  141.92  611.84  140.93  634.47   141.1 668.903  143.04
 688.982  142.78 702.138  140.32 727.281  140.49 760.301   142.9  811.54   143.1
 862.131  142.53 972.861  142.241024.236  141.811074.019  142.22 1089.11  144.37
 1117.39   147.1 1163.93  149.71 1217.36  151.82 1241.42  152.44 1279.22  152.24
IW Dist,WD,Coef,Skew,MaxSub,Min_El,Is_Ogee,SpillHt,DesHd
31.7,8,2.6,0,0.98,, 0 ,,,2,5,

Type RM Length L Ch R = 1 ,5222    ,400.13,476.37,422.46
XS GIS Cut Line= 3
 2301662.8313402  736752.1778436 2301101.8224662  736847.2914171
 2300750.9575375  736989.9389106
#Sta/Elev= 30
       0  147.73   27.39  146.59    63.6   145.7  103.83  143.52  172.56  141.47
  256.84  139.46  300.14  140.06  321.58  139.47  348.39  137.16  387.83  135.82
  407.98  135.63  429.24  133.66  440.15  132.46  447.83  132.82  452.59  133.66
  455.28  134.15  503.99  136.16  525.61  136.33  545.06  137.58  550.75  137.54
  580.44  137.61  608.93  138.39  636.27  137.77  647.21   137.1  660.04  137.37
  710.54  140.92  734.75  141.87  808.45  143.59   906.5  148.45  947.77  149.98
#Mann= 5 ,-1 , 0
       0    .045       0  387.83     .07       0  429.24     .05       0
  452.59     .08       0  550.75    .045       0
#XS Ineff= 2 , 0
       0                     615       0     141
Permanent Ineff=
       F       F
Bank Sta=429.24,452.59
XS Rating Curve= 0 ,0
Exp/Cntr=0.5,0.3

Type RM Length L Ch R = 1 ,4746    ,413.7,409.89,333.78
XS GIS Cut Line= 2
  2301610.375387  736375.0106218 2300681.8089749  736478.7334657
#Sta/Elev= 30
       0  148.04   34.34  146.83  114.59  143.22  143.55  142.75   193.1  140.85
   205.4  140.81  241.65  139.76  288.93  136.24  306.56  135.41  321.29  135.03
  333.02  135.22  354.58  132.94  365.67  131.82  377.19  132.84  408.43   135.4
  415.91   135.2  437.91  135.68     463  137.67  474.65  137.98   509.4  138.77
  551.86  140.93     588  143.85  627.17  146.19  639.88  146.64  652.95  146.59
  681.09  147.74   700.5  148.06  759.54  148.09  848.39  149.43  934.34  149.28
#Mann= 5 ,-1 , 0
       0    .045       0  306.56     .07       0  354.58     .05       0
  377.19     .08       0  474.65    .045       0
Bank Sta=354.58,377.19
XS Rating Curve= 0 ,0
Exp/Cntr=0.3,0.1

Type RM Length L Ch R = 1 ,4336    ,447.44,439.65,365.32
XS GIS Cut Line= 3
 2301526.4092753  735868.7443599 2300999.3718549  736123.6513475
  2300810.227734   736394.767354
#Sta/Elev= 30
       0  148.69   25.83   148.6   80.64  147.36  109.24  146.29  140.46  143.06
  150.11  141.01   159.2  140.29  197.12  139.83  240.66  136.73  251.14  136.42
  277.11  136.25  348.14  134.18  398.19   134.7  424.15  134.36  428.63  134.27
  434.51  132.84  440.33  131.43   458.1  132.85  479.59  134.75  499.04  135.36
   522.2  137.56  551.37  138.16  585.45  139.83  600.01   140.1  655.04  143.11
   719.9  145.09  735.95  145.62  777.93  145.41  882.18  148.24  916.02   148.8
#Mann= 5 ,-1 , 0
       0    .045       0   159.2     .07       0  434.51     .05       0
   458.1     .08       0   719.9    .045       0
Bank Sta=434.51,458.1
XS Rating Curve= 0 ,0
Exp/Cntr=0.3,0.1

Type RM Length L Ch R = 1 ,3896    ,399.59,404.36,413.44
XS GIS Cut Line= 3
  2301217.710335   735589.680518  2300923.828944   735703.281728
 2300543.5118497   736110.764329
#Sta/Elev= 30
       0  143.72   36.12  143.66   46.75  143.23  119.26   142.9  203.84  141.88
  327.48  137.78  366.93   137.1  390.09  135.63  393.92  135.61  412.39  135.54
   417.1  134.42  427.31  133.47  440.69  133.63  442.82  132.72  444.52  132.47
  455.75  130.79  463.48  132.45  464.77  132.88  500.11  136.32  534.22  137.54
  544.43  139.03  589.86  138.96  595.34  139.46  612.38  138.49  617.74  138.22
  639.85  138.71  658.65  139.52  706.63   140.2  815.94  144.35  872.46  145.94
#Mann= 5 ,-1 , 0
       0    .045       0  393.92     .07       0  444.52     .05       0
  463.48     .08       0  612.38    .045       0
#XS Ineff= 2 , 0
       0                     528       0     139
Permanent Ineff=
       F       F
Bank Sta=444.52,463.48
XS Rating Curve= 0 ,0
Exp/Cntr=0.3,0.1

Type RM Length L Ch R = 1 ,3492    ,510.28,509.35,505.53
XS GIS Cut Line= 2
 2300763.3054951  735315.5558591 2300259.5088247  735794.6566143
#Sta/Elev= 30
       0  144.27   20.19  143.65   40.56  142.73   63.58  141.42  110.23  139.61
  162.14  138.43  179.03  138.34  194.67     136  202.45  134.86  216.04  133.84
  237.86  133.58  247.06   133.1  262.36  133.04  282.74  133.41  292.07  133.36
  303.16  132.82  314.52  133.17  325.84  131.44  333.03  130.07  340.91  131.44
  347.76  132.51  352.28  132.69  411.09  133.99  427.94  134.38   466.5137.4501
  503.89   138.4  541.17  138.94  559.58  139.43  599.39  140.61  695.23  143.96
#Mann= 6 ,-1 , 0
       0    .045       0  194.67     .07       0  325.84     .05       0
  340.91     .08       0  411.09    .085       0   466.5    .045       0
Bank Sta=325.84,340.91
XS Rating Curve= 0 ,0
Exp/Cntr=0.3,0.1

Type RM Length L Ch R = 1 ,2983    ,506.74,506.11,515.51
XS GIS Cut Line= 2
 2300531.1638921  734831.5159209 2299896.4788711  735446.4442098
#Sta/Elev= 30
       0  139.55   34.97  138.76   55.71  139.81  116.09  139.87  166.52  139.38
  212.13  138.55  279.68  135.53  289.42  135.53  312.54  135.24  347.96  133.57
   388.1  132.82  412.53  132.81  447.73  133.22  480.25  129.93  496.75  128.28
  506.55  129.95  514.61  131.32  556.94   132.4  569.86  132.37  573.09  132.14
  581.21  131.69  606.25  132.33  647.42  134.26  657.84  134.38  696.46  134.72
  745.09  136.33  809.13   138.8   853.7  141.11  876.09   141.5  883.72  143.02
#Mann= 6 ,-1 , 0
       0    .045       0  289.42    .085       0  480.25     .05       0
  506.55     .08       0  573.09    .085       0  657.84    .045       0
Bank Sta=480.25,506.55
XS Rating Curve= 0 ,0
Exp/Cntr=0.3,0.1

Type RM Length L Ch R = 1 ,2476    ,125.56,150.05,196.92
XS GIS Cut Line= 4
 2300004.3053852  734730.3492017 2299846.3047714  734800.8802058
 2299800.0939023  734835.8376508 2299502.0088758  735061.3320231
#Sta/Elev= 30
       0  141.46   11.25  141.25   23.55  141.58   54.31  140.44   67.62  138.82
   77.74  138.68   87.65  137.63   95.07  137.32   150.9  134.61  166.85  134.02
  179.33  133.37  183.69  132.02  193.78  128.02  196.74  126.82  202.86  126.93
  214.39  128.01   240.1  130.44  278.66  131.23  280.65  131.45  294.09  131.47
  324.79  132.05  362.53  133.95  377.97  134.39  393.04  135.33  420.37  136.27
  430.98  136.95  442.06  138.22  466.68  138.64  532.85  142.22  604.74  143.82
#Mann= 6 ,-1 , 0
       0     .05       0   95.07    .045       0  166.85    .085       0
  193.78     .05       0  214.39    .085       0  294.09    .045       0
#XS Ineff= 2 , 0
       0   31.83  151.46               0
Permanent Ineff=
       F       F
#Block Obstruct= 1 ,-1
       0   31.83 151.462
Bank Sta=193.78,214.39
XS Rating Curve= 0 ,0
Exp/Cntr=0.5,0.3

Type RM Length L Ch R = 1 ,2326    ,70.46,65.43,58.23
BEGIN DESCRIPTION:
Surveyed Section
END DESCRIPTION:
XS GIS Cut Line= 6
 2299998.1692327  734650.6391228  2299798.574519  734699.3976698
    2299778.0333      734694.917    2299741.0911     734699.2527
    2299677.1594     734714.5897 2299397.4378096  734825.0690048
#Sta/Elev= 30
       0  142.24   40.49  140.98   71.34  139.78  107.02  139.06  118.58  139.15
  123.77  138.99  136.69  137.23  158.43  135.48  174.34  133.78  190.22  132.96
  225.39  132.06 226.329  131.85 256.645  129.66  260.69  128.09 263.612  126.94
 265.698  126.76 268.803  127.13  272.09  128.07 279.968  130.44  287.65  130.61
  346.62  132.03  387.74  132.46  405.78  132.97  434.55  133.45  473.79  133.41
     492  136.15  506.97  136.08  563.71  137.99  614.47  140.96  631.44  142.15
#Mann= 4 ,-1 , 0
       0     .05       0  260.69     .05       0  272.09    .085       0
  287.65    .045       0
#XS Ineff= 3 ,-1
       0   32.17  152.24   32.17  251.75  132.38  281.25     700   131.6
Permanent Ineff=
       F       F       F
#Block Obstruct= 1 ,-1
       0   32.17 152.236
Bank Sta=260.69,272.09
XS Rating Curve= 0 ,0
Exp/Cntr=0.5,0.3

Type RM Length L Ch R = 2 ,2300    ,,,
Node Photo=..\..\..\..\SURVEY\DTL\Surveys\Wilson\Bloomery Swamp Tributary 3\STR_34\STR_34 Photos\STR_34PHT2.JPG
Bridge Culvert--1,0,-1,-1, 0
Deck Dist Width WeirC Skew NumUp NumDn MinLoCord MaxHiCord MaxSubmerge Is_Ogee
21.2,10.1,2.6,0, 36, 36, , , 0.98, 0, 0,0,,
       0    7.61   14.37   22.42   29.93    72.6  109.13  144.52  148.05  161.96
  164.25  175.65 193.675 221.629 252.975 280.403 325.247  354.83  412.56  455.89
  459.05  483.01     504  525.19  542.72  549.77  564.11  567.76  579.23  590.69
  592.71  594.72  605.04  612.85  620.07  631.44
  141.89  141.66  141.47   141.2  140.92  139.64  139.12  136.47  136.24  134.65
  134.29   133.2  132.82  132.46  132.38  132.18   131.6  131.93  132.31  133.01
  133.04  134.76  136.53  136.49  137.17  137.53  138.33  138.54  139.22  139.59
  139.67  139.77  140.28  140.72  141.07  141.53
                                                                                
                                                                                
                                                                                
                                                
       0    7.61   14.37   22.42   29.93    72.6  109.13  144.52  148.05  161.96
  164.25  175.65 193.675 221.629 252.975 280.403 325.247  354.83  412.56  455.89
  459.05  483.01     504  525.19  542.72  549.77  564.11  567.76  579.23  590.69
  592.71  594.72  605.04  612.85  620.07  631.44
  141.89  141.66  141.47   141.2  140.92  139.64  139.12  136.47  136.24  134.65
  134.29   133.2  132.82  132.46  132.38  132.18   131.6  131.93  132.31  133.01
  133.04  134.76  136.53  136.49  137.17  137.53  138.33  138.54  139.22  139.59
  139.67  139.77  140.28  140.72  141.07  141.53
                                                                                
                                                                                
                                                                                
                                                
BR Coef=-1 , 0 , 0 ,, 0 ,,,0.8,-1,,0,
WSPro=,,,, 1 ,,,, 0 ,,,, 0 ,,,,-1 ,-1 ,-1 , 0 , 0 , 0 , 0 , 0
Multiple Barrel Culv=1,2,,21,0.012,0.5,1,1,1,126.11,126.4, 4,Culvert #3  , 0 ,14.9
  262.75  260.75  265.25  263.25  267.75  265.75  270.25  268.25
Culvert Bottom n=0.012
Culvert Bottom Depth=2
Culvert Depth Blocked=1.99
Culvert=1,2,,21,0.012,0.5,1,1,1,128.45,263.5,128.74,261.5,Culvert #1  , 0 ,14.9
Culvert Bottom n=0.012
Culvert Bottom Depth=2
Culvert Depth Blocked=1.5
Culvert=1,2,,21,0.012,0.5,1,1,1,128.45,266,128.74,264,Culvert #2  , 0 ,14.9
Culvert Bottom n=0.012
BC Design=,, 0 ,, 0 ,,,,,,
BC Use User HTab Curves=0
BC User HTab FreeFlow(D)= 0

Type RM Length L Ch R = 1 ,2261    ,170.6,177.05,176.14
BEGIN DESCRIPTION:
Surveyed Section
END DESCRIPTION:
XS GIS Cut Line= 6
 2299961.8445074   734578.538426 2299765.4450589  734635.3174136
    2299717.4365     734634.0792    2299703.1458     734654.1132
 2299659.4765283  734658.0442131 2299376.0173797  734773.0820108
#Sta/Elev= 30
       0  142.48   45.01  141.27    60.5  141.03   86.23  140.24   127.3  138.76
  137.28  138.17  154.27  137.74  195.09  134.22  206.92  133.49  235.07   132.6
 252.373  132.31 257.165  127.96 262.405  126.88 265.447  126.68  268.65   126.8
  271.67  127.97 277.371  130.23  301.63  130.21  338.56  131.38  349.24  131.94
  369.64   132.3  431.83  132.09  456.85   132.6   461.3  132.79  478.89  135.29
   499.5  136.59   521.3   136.4  535.59  136.83  593.95  139.68  627.23  140.99
#Mann= 4 ,-1 , 0
       0    .045       0 257.165     .05       0  271.67    .075       0
  349.24    .045       0
#XS Ineff= 3 ,-1
       0   79.33  151.35   79.33  249.75  130.74  279.25     700  130.74
Permanent Ineff=
       F       F       F
#Block Obstruct= 1 ,-1
   30.22   79.33 151.346
Bank Sta=257.165,271.67
XS Rating Curve= 0 ,0
Exp/Cntr=0.5,0.3

Type RM Length L Ch R = 1 ,2084    ,219.37,233.35,248.1
XS GIS Cut Line= 4
  2299814.865779  734469.3190467 2299668.4789635  734484.6927535
 2299506.7596575  734529.5544849 2299263.0678564  734630.1224333
#Sta/Elev= 30
       0   140.7   20.38  139.66   43.24  139.08   47.74  138.43   57.51  137.45
   81.62  136.28      96  135.18  105.78  134.66  152.71  131.01  175.27  129.53
  190.74  125.72  197.23  124.12  203.58  125.73   215.8  128.84  220.19  129.02
  242.69  128.08  287.43  128.67  315.29  129.49  331.59  129.73  339.13  130.12
  353.28   130.2  362.66  130.73  417.86  132.61  439.34  133.72  485.74  135.56
   501.9  136.39  542.67  137.71  565.45  138.83  572.79  139.66  578.65  139.99
#Mann= 4 ,-1 , 0
       0    .045       0  190.74     .05       0   215.8    .075       0
  565.45    .045       0
#XS Ineff= 2 , 0
       0                     340       0
Permanent Ineff=
       F       F
Bank Sta=190.74,203.58
XS Rating Curve= 0 ,0
Exp/Cntr=0.3,0.1

Type RM Length L Ch R = 1 ,1851    ,137.65,142.7,129.08
XS GIS Cut Line= 3
 2299892.2276823  734268.4516211 2299653.9300705  734265.9563582
 2299207.2780023  734313.3663543
#Sta/Elev= 30
       0  141.25   30.82  140.59   39.43   139.5   51.33  138.42   76.81  136.93
  117.52  134.99  138.47  134.64  151.44   133.8  159.67  132.57  177.73  131.85
  203.52  130.21  279.34  127.32  293.12  127.25  310.35  126.73  320.35  124.76
  328.18  122.89  335.52  124.93  349.69  126.83  353.56   127.1  367.66   126.9
   380.2  127.26  425.05  127.72  469.56  129.11  491.89  130.49  536.67  133.83
  554.99  135.44  572.59  136.46  609.34  137.72  651.87  138.61  687.47  138.95
#Mann= 3 , 0 , 0
       0    .045       0  320.35     .05       0  335.52    .075       0
#XS Ineff= 2 , 0
       0     200             450       0
Permanent Ineff=
       F       F
Bank Sta=320.35,335.52
XS Rating Curve= 0 ,0
Exp/Cntr=0.5,0.3

Type RM Length L Ch R = 1 ,1708    ,245.72,230.83,210.96
BEGIN DESCRIPTION:
Surveyed Section
END DESCRIPTION:
XS GIS Cut Line= 6
 2300346.1992795  733766.7514361 2299740.0166423   734095.030846
    2299607.2487     734140.4808     2299500.758     734146.5554
 2299335.7840443  734186.1079438 2299053.8193308  734212.3082047
#Sta/Elev= 30
       0  139.37   13.06  139.19  168.12138.1551  220.73  137.66  236.91  137.04
  294.17  137.87  345.82  137.44  398.64  136.74  417.28  135.71  469.43  137.16
  509.43  137.19  549.56   136.6  635.76  133.83  722.45  130.35  826.34  127.59
 875.146  126.85 886.597  124.39 889.728  122.75  892.16  122.26 895.065  122.73
  898.06   124.4 902.562  126.94 936.466  127.44  950.83  128.23  976.03  128.18
 1021.67  129.27 1066.88  132.64 1122.46  135.73  1261.1  138.13 1389.38  139.12
#Mann= 6 ,-1 , 0
       0     .03       0   13.06    .045       0  168.12    .055       0
  345.82    .045       0 886.597     .05       0  898.06    .075       0
#XS Ineff= 3 ,-1
       0  282.89  147.63  282.89     869  133.05     911    1400  134.07
Permanent Ineff=
       F       F       F
#Block Obstruct= 1 ,-1
  234.81  282.89 147.635
Bank Sta=886.597,898.06
XS Rating Curve= 0 ,0
Exp/Cntr=0.5,0.3

Type RM Length L Ch R = 2 ,1613    ,,,
BEGIN DESCRIPTION:
Raleigh Road (264 Bus.)
END DESCRIPTION:
Bridge Culvert--1,0,-1,-1, 0
Deck Dist Width WeirC Skew NumUp NumDn MinLoCord MaxHiCord MaxSubmerge Is_Ogee
75.8,101.5,2.6,0, 18, 17, , , 0.98, 0, 1,1,,
       0    23.1  214.89  393.83  516.02  606.71 750.955 834.479 875.301 916.401
 998.446 1079.57 1154.54 1265.78 1329.29 1376.31 1387.36 1389.38
  138.04  137.89  136.26  134.86  133.93  133.46  133.05  133.42  133.79  134.17
  135.22  136.79  137.96  139.54  140.71   141.3   141.3   141.3
                                                                                
                                                                
       0    23.1  214.89  393.83  516.02  606.71 750.955 834.479 875.301 916.401
 998.446 1079.57 1154.54 1265.78 1329.29 1376.31 1387.36
  138.04  137.89  136.26  134.86  133.93  133.46  133.05  133.42  133.79  134.17
  135.22  136.79  137.96  139.54  140.71   141.3   141.3
                                                                                
                                                        
BR Coef=-1 , 0 , 0 ,, 0 ,,,0.8,-1,,0,
WSPro=,,,, 1 ,,,, 0 ,,,, 0 ,,,,-1 ,-1 ,-1 , 0 , 0 , 0 , 0 , 0
Multiple Barrel Culv=2,6,6,142.7,0.011,0.4,1,8,1,122.04,120.63, 2,Culvert #1  , 0 ,47
  886.75  868.75  893.25  875.25
Culvert Bottom n=0.011
BC Design=,, 0 ,, 0 ,,,,,,
BC Use User HTab Curves=0
BC User HTab FreeFlow(D)= 0

Type RM Length L Ch R = 1 ,1477    ,161.1,193.44,201.43
BEGIN DESCRIPTION:
Surveyed Section
END DESCRIPTION:
XS GIS Cut Line= 6
 2300297.7079119  733527.3585247 2299758.7311145    733819.30429
 2299663.9111223  733862.9713916    2299449.2396     733943.9731
 2299322.0600981  733974.0105929 2299067.5432771  733998.9632224
#Sta/Elev= 30
       0  138.15   36.93  137.27   57.24  135.86   99.59  134.35  249.46  131.88
  423.06  130.34  451.05   130.8  467.01  130.14   473.1  131.71   520.6  131.56
  624.68  132.34  644.66  131.28  682.16  130.55  723.79  128.38  794.63  126.67
  805.09  125.71  853.61 126.301 859.316  126.37  863.78  123.91 866.361  122.44
 873.671  120.72 881.029   123.9 891.672  128.16 947.434  129.66 1082.22  134.56
 1147.78  135.28 1156.92  135.88 1181.92  135.27 1217.44  136.29 1334.18  136.46
#Mann= 6 ,-1 , 0
       0     .04       0   473.1    .055       0  723.79    .075       0
  853.61    .085       0  863.78     .05       0 881.029     .05       0
#XS Ineff= 2 ,-1
       0     850  133.05  888.25    1400  133.91
Permanent Ineff=
       F       F
Bank Sta=863.78,881.029
XS Rating Curve= 0 ,0
Exp/Cntr=0.5,0.3

Type RM Length L Ch R = 1 ,1284    ,323.12,452.16,364.1
XS GIS Cut Line= 4
 2300121.7918739  733468.8757993 2299604.0248115  733726.1997911
 2299323.3077295  733765.1882747 2299069.1028164  733882.1537256
#Sta/Elev= 30
       0  133.77   90.68  131.44  170.58  130.07  279.75  128.75  312.93  129.18
  323.02  128.65  344.23  129.81  365.66  130.29  397.12  130.02  416.67  129.37
  472.87  129.29  507.35  127.46  537.72  126.95   656.2  125.02  726.25  125.99
  742.93   123.9  750.37  122.49  760.02  121.08   763.4  122.46  767.16  124.05
  775.22  125.72  785.18  126.54  791.73  127.05  811.26  126.93  817.63  127.32
  881.03  128.11  958.36  130.41   997.4   130.7 1017.48  132.13 1141.42  133.95
#Mann= 7 ,-1 , 0
       0     .04       0  323.02    .055       0  537.72    .075       0
   656.2    .085       0  750.37     .05       0   763.4    .085       0
  785.18     .05       0
#XS Ineff= 2 ,-1
       0  464.04   139.6  464.04     630     129
Permanent Ineff=
       F       F
#Block Obstruct= 2 ,-1
  332.86  353.77 140.052  430.04  464.04 139.599
Bank Sta=750.37,763.4
XS Rating Curve= 0 ,0
Exp/Cntr=0.3,0.1

Type RM Length L Ch R = 1 ,831     ,259.2,253.54,183.08
XS GIS Cut Line= 3
 2299866.0274213  733375.3034386 2299658.6086886  733411.1728435
 2299187.6278065   733386.220214
#Sta/Elev= 30
       0  131.48   51.03  131.02   82.88  129.74   87.11  129.84  115.28  130.75
  125.35  129.96  134.14  128.36  150.32  127.78  155.86  127.03  171.33  127.12
  184.85  128.28   211.7  127.01  218.99  126.02  241.99  121.97  247.41  121.02
  256.11  121.97   316.8  124.79  342.54  123.56  358.66  123.89  380.67   124.9
  421.14  124.67  430.02  124.37  433.92  124.32  463.96  126.26  513.06  127.58
  527.08  128.12  552.37   129.8  594.85  131.17  650.75  131.86  682.14  131.74
#Mann= 5 ,-1 , 0
       0     .04       0   87.11    .085       0  241.99     .05       0
  256.11    .085       0  430.02     .05       0
#XS Ineff= 2 , 0
       0  184.85  128.28     342       0
Permanent Ineff=
       F       F
Bank Sta=241.99,256.11
XS Rating Curve= 0 ,0
Exp/Cntr=0.3,0.1

Type RM Length L Ch R = 1 ,578     ,339.27,344.68,257.07
XS GIS Cut Line= 2
 2299716.3116443  733133.5748403 2299162.6751771  733323.8386403
#Sta/Elev= 30
       0  136.95   13.84  136.47   19.79  136.58   32.12  136.03   55.73  133.13
   67.25  125.63   74.26  122.14   76.52  120.99   79.41  122.14   88.46  124.16
  110.83  126.26  117.66  125.53  139.94  124.86  182.23  122.77  237.29  122.23
  252.39  122.59  272.75  121.27  276.82  121.69  283.01  121.61  287.62  121.93
   327.1  125.23  365.65  126.59  411.66  128.81  496.24  130.75  503.38  130.14
  540.62  130.37  543.06  130.66  562.89  131.02  571.56  131.76  585.16  132.04
#Mann= 5 ,-1 , 0
       0     .04       0   19.79    .085       0   74.26     .05       0
   79.41    .085       0  287.62     .05       0
#XS Ineff= 2 , 0
       0                     220       0
Permanent Ineff=
       F       F
Bank Sta=74.26,79.41
XS Rating Curve= 0 ,0
Exp/Cntr=0.3,0.1

Type RM Length L Ch R = 1 ,233     ,158.26,175.14,106.72
XS GIS Cut Line= 4
 2299608.7034296  732801.3929599 2299507.3333722  732851.2982189
 2299348.4070689  733003.4683942  2299148.639323  733298.8860108
#Sta/Elev= 30
       0  133.56    8.96  133.69   17.93  133.29      27  132.92   46.84  132.67
   77.32   130.9  108.69  130.27     148  121.21   152.8  120.08  164.13  121.19
  189.38  124.11  192.47  123.98  205.38  122.07  228.19  121.48  271.85  121.15
  320.51  122.27  326.34  121.38  330.42  120.75   331.9  121.02  332.56  120.75
   401.4  125.51  412.42  126.53  429.35  127.39  459.89  127.83  518.54  129.59
  583.45  130.26  601.79  129.94  632.63  131.25  645.03  131.24  689.54  132.01
#Mann= 5 ,-1 , 0
       0     .04       0   17.93    .085       0     148     .05       0
  164.13    .085       0  326.34     .05       0
#XS Ineff= 1 ,-1
     290     700  136.63
Permanent Ineff=
       F
#Block Obstruct= 1 ,-1
  349.97  414.37 136.628
Bank Sta=148,164.13
XS Rating Curve= 0 ,0
Exp/Cntr=0.3,0.1
