HEC-RAS study Town_Creek_FINAL.prj: Town Creek

--- Town_Creek_FINAL.g01 (geometry) --- (continued)

Type RM Length L Ch R = 1 ,157006.3,501.2,501.2,501.2
BEGIN DESCRIPTION:
Town Creek 312.0
END DESCRIPTION:
#Sta/Elev= 26
  4192.4  103.72  4292.4    94.9  4332.4   88.82  4432.4   79.86  4452.4   79.08
  4462.4   78.02  4492.4   76.97  4522.4   78.74  4572.4   78.72  4592.4   77.71
  4632.4   79.05  4842.4    78.1  4942.4   79.22  4982.2   76.38  4983.7   73.38
  5016.3   73.38  5017.8   76.38    5050   78.81    5140   78.17    5180   79.65
    5340   80.48    6040   82.11    6180   81.73    6350   88.67    6390   93.95
  6426.9   97.29
#Mann= 3 , 1 , 0
 4192.40   0.135       0  4982.2    0.05       0  5017.8   0.135       0
Bank Sta=4982.20,5017.80
Exp/Cntr=0.3,0.1

Type RM Length L Ch R = 1 ,156505.1,498.1,498.1,498.1
BEGIN DESCRIPTION:
Town Creek 311.0
END DESCRIPTION:
#Sta/Elev= 30
  4236.7   97.98  4276.7   92.91  4306.7    87.7  4346.7   83.28  4406.7   81.63
  4456.7   78.13  4636.7   77.22  4686.7   78.38  4766.7   78.27  4806.7   76.43
  4966.7   77.35  4982.2   76.03  4983.7   73.03  5016.3   73.03  5017.8   76.03
    5040   75.94    5080   77.39    5220   76.95  5279.8   78.02  5419.8   77.79
  5489.8   77.25  5529.8   80.76  5559.8   81.65  5599.8    81.6  5609.8   81.05
  5669.8   82.77  5709.8   82.97  5752.1   82.85    5870   83.62  5892.1   83.76
#Mann= 4 , 1 , 0
 4236.70   0.135       0  4982.2    0.05       0  5017.8   0.135       0
    5870    0.18       0
Bank Sta=4982.20,5017.80
Exp/Cntr=0.3,0.1

Type RM Length L Ch R = 1 ,156007.0,600.2,600.2,600.2
BEGIN DESCRIPTION:
Town Creek 310.0
END DESCRIPTION:
#Sta/Elev= 24
  4382.5   96.84  4512.5   88.14  4602.5   84.53  4682.5   77.21  4722.5    76.2
  4742.5   76.43  4802.5   75.81  4862.5   76.77  4912.5   75.96  4982.1   75.68
  4983.6   72.68  5016.3   72.68  5017.8   75.68    5040   76.75    5110   76.31
    5190   76.72    5410   76.58    5460   75.97    5640    76.4    5660   75.89
    5730   76.74    5810   84.87    5870   88.74  5927.2   91.79
#Mann= 3 , 1 , 0
 4382.50   0.135       0  4982.1    0.05       0  5017.8   0.135       0
Bank Sta=4982.10,5017.80
Exp/Cntr=0.3,0.1

Type RM Length L Ch R = 1 ,155406.8,571.5,571.5,571.5
BEGIN DESCRIPTION:
Town Creek 309.0
END DESCRIPTION:
#Sta/Elev= 26
  4452.9   92.14  4492.9   91.76  4502.9   92.37  4522.9   91.23  4532.9   91.53
  4542.9   92.71  4552.9   93.22  4562.9   91.92  4582.9    90.8  4592.9   89.82
  4662.9   86.41  4732.9   84.87  4812.9   82.62  4882.9    80.9  4932.9   77.59
  4982.2   75.25  4983.7   72.25  5016.3   72.25  5017.8   75.25  5506.4   75.28
  5576.4   76.01  5676.4   75.26  5696.4   76.14  5736.4   82.08  5846.4    92.2
    5936   97.79
#Mann= 3 , 1 , 0
 4452.90   0.135       0  4982.2    0.05       0  5017.8   0.135       0
Bank Sta=4982.20,5017.80
Exp/Cntr=0.3,0.1

Type RM Length L Ch R = 1 ,154835.3,688.4,688.4,688.4
BEGIN DESCRIPTION:
Town Creek 308.0
END DESCRIPTION:
#Sta/Elev= 30
  4143.9   93.06  4163.9   91.47  4403.9   84.98  4413.9   85.01  4433.9    86.9
  4453.9   83.18  4553.9   80.43  4623.9   75.32  4643.9   75.45  4663.9   76.71
  4733.9   77.64  4823.9   76.07  4863.9   76.65  4873.9   76.02  4903.9   76.39
  4982.2   74.85  4983.7   71.85  5016.3   71.85  5017.8   74.85  5110.5    74.9
  5190.5   74.72  5210.5   75.47  5310.5    76.2  5370.5   80.37  5380.5   80.36
  5420.5   82.65  5450.5   85.04  5580.5   89.18  5740.5  101.32    5773  102.72
#Mann= 3 , 1 , 0
 4143.90   0.135       0  4982.2    0.05       0  5017.8   0.135       0
Bank Sta=4982.20,5017.80
Exp/Cntr=0.3,0.1

Type RM Length L Ch R = 1 ,154146.9,633.8,633.8,633.8
BEGIN DESCRIPTION:
Town Creek 306.0
END DESCRIPTION:
#Sta/Elev= 30
  3753.4   92.11  3883.4   85.43  3923.4   84.58  3973.4   81.85  3983.4   80.55
  3993.4   80.15  4223.8   81.27  4513.8   80.93  4623.8   76.09  4643.8   75.79
  4793.8   75.92  4953.8   74.45  4980.7   75.03  4982.2   74.36  4983.7   71.36
  5016.4   71.36  5017.9   74.36  5030.7   75.42  5150.7   74.78  5170.7   76.18
  5210.7   82.62  5240.7   82.71  5260.7   83.89  5290.7   83.81  5300.7   84.74
  5320.7    85.1  5360.7   84.44  5470.7   85.79  5570.7   89.23  5642.3   95.31
#Mann= 3 , 1 , 0
 3753.40   0.135       0  4982.2    0.05       0  5017.9   0.135       0
Bank Sta=4982.20,5017.90
Exp/Cntr=0.3,0.1

Type RM Length L Ch R = 1 ,153513.1,578.5,578.5,578.5
BEGIN DESCRIPTION:
Town Creek 305.0
END DESCRIPTION:
#Sta/Elev= 24
  3299.8   89.85  3429.8   82.77  3479.8   77.98  3489.8   78.54  3499.8    79.6
  4417.6   79.54  4447.6    80.1  4567.6   79.25  4607.6   75.55  4757.6   75.67
  4982.2   73.92  4983.7   70.92  5016.3   70.92  5017.8   73.92    5070   75.17
    5180   74.57    5270   75.31    5280   75.77    5290   76.79    5310   80.43
    5330   84.99    5350   90.36    5360   92.62  5361.1   92.83
#Mann= 3 , 1 , 0
 3299.80   0.135       0  4982.2    0.05       0  5017.8   0.135       0
Bank Sta=4982.20,5017.80
Exp/Cntr=0.3,0.1

Type RM Length L Ch R = 1 ,152934.6,917.1,917.1,917.1
BEGIN DESCRIPTION:
Town Creek 304.0
END DESCRIPTION:
#Sta/Elev= 26
  3011.8   90.61  3151.8   81.48  4041.8   81.99  4051.8   82.39  4451.8   79.17
  4501.8   75.74  4581.8    75.6  4661.8   76.43  4701.8   80.16  4791.6   80.58
  4871.6   78.58  4901.6   76.62  4971.6   76.07  4981.6   75.47  4982.2   73.51
  4983.7   70.51  5016.3   70.51  5017.8   73.51  5021.6   75.59  5173.7    75.2
  5333.7   74.86  5343.7   76.75  5363.7   82.65  5373.7   85.13  5383.7   87.09
  5425.1   92.49
#Mann= 3 , 1 , 0
 3011.80   0.135       0  4982.2    0.05       0  5017.8   0.135       0
Bank Sta=4982.20,5017.80
Exp/Cntr=0.3,0.1

Type RM Length L Ch R = 1 ,152017.5,499.5,499.5,499.5
BEGIN DESCRIPTION:
Town Creek 302.0
END DESCRIPTION:
#Sta/Elev= 30
  2511.6   89.06  2621.6   81.79  3531.6   81.49  3551.6   81.81  3991.6   79.09
  4161.6   79.94  4181.6   78.55  4191.6   77.45  4421.6    79.2    4459    78.3
    4499   77.83    4599   78.18    4629   77.28    4669   77.38    4709   78.05
    4739    77.6    4949   75.17  4982.2   72.86  4983.7   69.86  5016.3   69.86
  5017.8   72.86    5140   75.28    5150   75.69    5160   76.69    5170   76.97
    5210   81.83    5220   83.66    5250   84.96    5400   85.96  5753.1   86.29
#Mann= 3 , 1 , 0
 2511.60   0.135       0  4982.2    0.05       0  5017.8   0.135       0
Bank Sta=4982.20,5017.80
Exp/Cntr=0.3,0.1

Type RM Length L Ch R = 1 ,151518.0,785.9,785.9,785.9
BEGIN DESCRIPTION:
Town Creek 301.0
END DESCRIPTION:
#Sta/Elev= 30
  2443.1   89.53  2553.1   82.06  2563.1   81.09  2583.1   80.85  2623.1   80.18
  3833.1   80.11  3869.6   80.31  3939.6   80.15  3959.6   79.08  4129.6   77.59
  4219.6   77.21  4239.6   76.81  4329.6    78.5  4479.6   76.43  4539.6   77.65
  4599.6   73.48  4659.6   74.46  4679.6   74.19  4969.2   72.51  4970.7   69.51
  5029.4   69.51  5030.9   72.51    5330   75.88    5390   78.85    5540   77.17
    5550   76.69    5620   80.26  5633.1    80.3  5933.1    84.2  6100.3   86.16
#Mann= 3 , 1 , 0
 2443.10   0.135       0  4969.2    0.05       0  5030.9   0.135       0
Bank Sta=4969.20,5030.90
Exp/Cntr=0.3,0.1

Type RM Length L Ch R = 1 ,150732.1,713.9,713.9,713.9
BEGIN DESCRIPTION:
Town Creek 299.0
END DESCRIPTION:
#Sta/Elev= 30
  2797.7   94.22  2877.7   87.56  2997.7   81.21  3017.7    80.8  3027.7   79.19
  3047.7   80.34  3227.7   80.94  4229.2   80.51  4329.2   80.56  4379.2   78.92
  4419.2   75.37  4439.2   75.45  4499.2   78.24  4569.2   77.68  4631.6   78.56
  4721.6   77.43  4751.6   77.68  4811.6   75.86  4851.6   72.92  4901.6   74.03
 4978.37   71.97 4979.42   68.97 5020.51   68.97 5021.56   71.97  5252.5   77.36
  5562.5   75.05  5702.5   77.31  5782.5   76.38  5802.5   78.05  5902.5   82.55
#Mann= 3 , 1 , 0
 2797.70   0.135       0 4978.37    0.05       0 5021.56   0.135       0
Bank Sta=4978.37,5021.56
Exp/Cntr=0.3,0.1

Type RM Length L Ch R = 1 ,150018.2,387,387,387
BEGIN DESCRIPTION:
Town Creek 298.0
END DESCRIPTION:
#Sta/Elev= 30
  3059.4   91.92  3949.4   79.38  4089.4   80.69  4139.4   78.14  4169.4   75.16
  4179.4   74.51  4209.4    76.5  4449.4   78.01  4539.4   75.35  4589.4   76.87
  4729.4   76.99  4749.4   77.49  4829.4    77.3  4909.4   72.63 4978.44   70.99
 4979.49   67.99 5020.58   67.99 5021.63   70.99    5130   76.23    5280   73.68
    5590   76.72    5670   76.41    5680   76.02    5760   78.13  6096.8   79.53
  6726.8   78.32  6736.8   78.99  6746.8   78.74  6766.8   80.57  6864.8   84.62
#Mann= 3 , 1 , 0
 3059.40   0.135       0 4978.44    0.05       0 5021.63   0.135       0
Bank Sta=4978.44,5021.63
Exp/Cntr=0.3,0.1

Type RM Length L Ch R = 1 ,149631.2,425.4,425.4,425.4
BEGIN DESCRIPTION:
Town Creek 297.0
END DESCRIPTION:
#Sta/Elev= 30
  3361.2    82.8  4276.6      80  4406.6      79  4436.6   76.81  4556.6   74.77
  4646.6    77.6  4786.6   76.52  4836.6   74.57  4946.6   74.79 4978.44   70.94
 4979.49   67.94 5020.51   67.94 5021.56   70.94  5036.1   73.53  5126.1   73.03
  5146.1   73.72  5176.1   73.33  5236.1   75.35  5346.1   73.28    5493    76.6
    5593   73.17  5862.9   78.77  6702.9   78.73  6722.9   78.01  6762.9   78.99
  6782.9   78.33  6792.9   81.65  6802.9   82.82  6832.9   83.25  6872.8   85.97
#Mann= 3 , 1 , 0
 3361.20   0.135       0 4978.44    0.05       0 5021.56   0.135       0
Bank Sta=4978.44,5021.56
Exp/Cntr=0.5,0.3

Type RM Length L Ch R = 1 ,149205.8,45,45,45
BEGIN DESCRIPTION:
Upstream Section of Bridge/Culvert/Weir
END DESCRIPTION:
#Sta/Elev= 30
  2786.8    89.5  3711.1   80.02  4391.2   78.79  4431.2   75.84  4560.4   76.83
  4590.4   76.04  4600.4   76.75  4767.6   76.09  4937.6   74.13  4976.5      73
    4980   67.91    5020   67.91  5023.5      73  5067.6   74.06    5108   72.87
    5198   72.66    5228   74.27    5298   74.95    5318   73.85    5408   74.99
  5663.6   74.28  5713.6   73.47  5793.6    74.2  5853.6   77.14  5943.6    74.9
  6083.6   77.57  6453.6    78.4  6543.6   79.83  6673.6    84.9  6701.7   86.63
#Mann= 3 , 1 , 0
 2786.80   0.135       0  4976.5    0.05       0  5023.5   0.135       0
#XS Ineff= 2 , 0
       0  4966.5   78.01  5033.5       0   76.83
Bank Sta=4976.50,5023.50
Exp/Cntr=0.5,0.3

Type RM Length L Ch R = 3 ,149183.3,,,
BEGIN DESCRIPTION:
Town Creek Road - TOR
Structure ID: Town Creek Road
Approximate Survey Structure
END DESCRIPTION:
Bridge Culvert--1,0,-1,-1, 0
Deck Dist Width WeirC Skew NumUp NumDn MinLoCord MaxHiCord MaxSubmerge Is_Ogee
10,25,2.6,, 60, 60,,,0.95,0,1,1,,
  2786.8  3625.3  3711.1  3805.3  3945.3  3983.2  4213.2  4311.2  4391.2  4431.2
  4460.4  4560.4  4590.4  4600.4  4717.6  4767.6  4937.6 4952.91    4953 5046.89
    5047  5067.6  5087.6    5108    5198    5228    5288    5298    5308    5318
    5408  5422.4  5542.4  5663.6  5713.6  5756.1  5793.6  5853.6  5943.6  5966.1
  5996.1  6016.1  6083.6  6126.1  6286.1  6336.1  6356.1  6403.6  6413.6  6453.6
  6466.1  6503.6  6513.6  6543.6  6573.6  6596.1  6623.9  6673.6  6693.6  6701.7
    89.5   80.91   80.26   80.29   80.02   79.65    78.8   78.94   78.85   78.69
   78.56   78.17   78.14   78.13   78.02   78.01   78.02   78.02   78.02      78
      78   77.97   77.94    77.9   77.72   77.66   77.54   77.52    77.5   77.48
   77.26   77.11   76.83   77.81   78.15   78.44   78.42   78.45   78.62   78.66
   79.15   78.73    78.7   79.33   79.38   80.97   81.04   80.65   80.51   79.99
   79.82   81.85   82.39   83.54   84.64   85.47   85.49   86.22   86.51   86.63
    89.5    80.9   80.02   79.79   79.45   79.36   78.79   78.47   78.79   75.84
    75.8   76.83   76.04   76.75   76.08   76.09   74.13   73.69   76.22    76.2
   73.56   74.06   73.63   72.87   72.66   74.27   74.58   74.95   73.98   73.85
   74.99   74.95   74.62   74.28   73.47   73.86    74.2   77.14    74.9   75.33
    75.9   76.28   77.57   77.68   78.02   78.06   78.08   78.11   78.55    78.4
   78.53   78.91   79.54   79.83   80.85   82.27   83.21    84.9   86.37   86.63
  2786.8  3625.3  3711.1  3805.3  3945.3  3983.2  4213.2  4311.2  4391.2  4431.2
  4460.4  4560.4  4590.4  4600.4  4717.6  4767.6  4937.6 4952.91    4953 5046.89
    5047  5067.6  5087.6    5108    5198    5228    5288    5298    5308    5318
    5408  5422.4  5542.4  5663.6  5713.6  5756.1  5793.6  5853.6  5943.6  5966.1
  5996.1  6016.1  6083.6  6126.1  6286.1  6336.1  6356.1  6403.6  6413.6  6453.6
  6466.1  6503.6  6513.6  6543.6  6573.6  6596.1  6623.9  6673.6  6693.6  6701.7
    89.5   80.91   80.26   80.29   80.02   79.65    78.8   78.94   78.85   78.69
   78.56   78.17   78.14   78.13   78.02   78.01   78.02   78.02   78.02      78
      78   77.97   77.94    77.9   77.72   77.66   77.54   77.52    77.5   77.48
   77.26   77.11   76.83   77.81   78.15   78.44   78.42   78.45   78.62   78.66
   79.15   78.73    78.7   79.33   79.38   80.97   81.04   80.65   80.51   79.99
   79.82   81.85   82.39   83.54   84.64   85.47   85.49   86.22   86.51   86.63
    89.5    80.9   80.02   79.79   79.45   79.36   78.79   78.47   78.79   75.84
    75.8   76.83   76.04   76.75   76.08   76.09   74.13   73.69   76.22    76.2
   73.56   74.06   73.63   72.87   72.66   74.27   74.58   74.95   73.98   73.85
   74.99   74.95   74.62   74.28   73.47   73.86    74.2   77.14    74.9   75.33
    75.9   76.28   77.57   77.68   78.02   78.06   78.08   78.11   78.55    78.4
   78.53   78.91   79.54   79.83   80.85   82.27   83.21    84.9   86.37   86.63
Pier Skew, UpSta & Num, DnSta & Num=,4968.0, 2 ,4968.0, 2 , 0 , 0 , 0 ,,
       1       1
   72.23   77.22
       1       1
   72.23   77.22
Pier Skew, UpSta & Num, DnSta & Num=,4984.0, 2 ,4984.0, 2 , 0 , 0 , 0 ,,
       1       1
   66.91   77.22
       1       1
   66.91   77.22
Pier Skew, UpSta & Num, DnSta & Num=,5000.0, 2 ,5000.0, 2 , 0 , 0 , 0 ,,
       1       1
   66.91   77.22
       1       1
   66.91   77.22
Pier Skew, UpSta & Num, DnSta & Num=,5016.0, 2 ,5016.0, 2 , 0 , 0 , 0 ,,
       1       1
   66.91   77.22
       1       1
   66.91   77.22
Pier Skew, UpSta & Num, DnSta & Num=,5032.0, 2 ,5032.0, 2 , 0 , 0 , 0 ,,
       1       1
    72.2   77.22
       1       1
    72.2   77.22
Abutment Skew #Up #Dn=, 2 , 2
 4952.80 4960.00
   76.22   73.48
 4952.80 4960.00
   76.22   73.48
Abutment Skew #Up #Dn=, 2 , 2
 5040.00 5047.09
   73.40   76.20
 5040.00 5047.09
   73.40   76.20
BR Coef= 1 , 1 , 0 ,1.25, 0 ,,,0.8,0,2,0,
Wspro=,,,, 1 ,,,, 0 ,,,, 0 ,,,,-1 ,-1 ,-1 , 0 , 0 , 0 , 0 , 0
BC Design=,, 0 ,, 0 ,,,,,,
BR U #Sta/Elev= 93
  2786.8    89.5  3335.3   83.87  3495.3   82.23  3515.3   82.03  3565.3   81.52
  3625.3    80.9  3711.1   80.02  3805.3   79.79  3945.3   79.45  3983.2   79.36
  4013.2   79.28  4073.2   79.14  4103.2   79.06  4183.2   78.87  4213.2   78.79
  4231.2   78.75  4311.2   78.47  4334.9   78.56  4391.2   78.79  4404.9   77.78
  4431.2   75.84  4460.4    75.8  4544.9   76.67  4560.4   76.83  4590.4   76.04
  4600.4   76.75  4717.6   76.08  4723.7   76.08  4767.6   76.09  4937.6   74.13
 4952.91   73.69    4953   73.68    4960   73.48  4976.5      73    4980   67.91
    5020   67.91  5023.5      73  5030.4   73.17    5040    73.4 5046.89   73.56
    5047   73.56  5067.6   74.06  5087.6   73.63  5100.4   73.15    5108   72.87
    5198   72.66    5228   74.27    5288   74.58    5298   74.95    5308   73.98
    5318   73.85  5336.4   74.08  5402.4   74.92    5408   74.99  5422.4   74.95
  5542.4   74.62  5582.4   74.51  5663.6   74.28  5713.6   73.47  5756.1   73.86
  5793.6    74.2  5826.1   75.79  5853.6   77.14  5943.6    74.9  5966.1   75.33
  5996.1    75.9  6016.1   76.28  6026.1   76.47  6083.6   77.57  6086.1   77.58
  6126.1   77.68  6166.1   77.78  6253.6      78  6286.1   78.02  6336.1   78.06
  6356.1   78.08  6396.1    78.1  6403.6   78.11  6413.6   78.55  6416.1   78.54
  6453.6    78.4  6466.1   78.53  6503.6   78.91  6513.6   79.54  6516.1   79.56
  6543.6   79.83  6573.6   80.85  6593.6   82.18  6596.1   82.27  6623.9   83.21
  6673.6    84.9  6693.6   86.37  6701.7   86.63
BR U #Mann= 3
 2786.80   0.135  4976.5    0.05  5023.5   0.135
BR U Banks=4976.50,5023.50
BR D #Sta/Elev= 93
  2786.8    89.5  3335.3   83.87  3495.3   82.23  3515.3   82.03  3565.3   81.52
  3625.3    80.9  3711.1   80.02  3805.3   79.79  3945.3   79.45  3983.2   79.36
  4013.2   79.28  4073.2   79.14  4103.2   79.06  4183.2   78.87  4213.2   78.79
  4231.2   78.75  4311.2   78.47  4334.9   78.56  4391.2   78.79  4404.9   77.78
  4431.2   75.84  4460.4    75.8  4544.9   76.67  4560.4   76.83  4590.4   76.04
  4600.4   76.75  4717.6   76.08  4723.7   76.08  4767.6   76.09  4937.6   74.13
 4952.91   73.69    4953   73.68    4960   73.48  4976.5      73    4980   67.91
    5020   67.91  5023.5      73  5030.4   73.17    5040    73.4 5046.89   73.56
    5047   73.56  5067.6   74.06  5087.6   73.63  5100.4   73.15    5108   72.87
    5198   72.66    5228   74.27    5288   74.58    5298   74.95    5308   73.98
    5318   73.85  5336.4   74.08  5402.4   74.92    5408   74.99  5422.4   74.95
  5542.4   74.62  5582.4   74.51  5663.6   74.28  5713.6   73.47  5756.1   73.86
  5793.6    74.2  5826.1   75.79  5853.6   77.14  5943.6    74.9  5966.1   75.33
  5996.1    75.9  6016.1   76.28  6026.1   76.47  6083.6   77.57  6086.1   77.58
  6126.1   77.68  6166.1   77.78  6253.6      78  6286.1   78.02  6336.1   78.06
  6356.1   78.08  6396.1    78.1  6403.6   78.11  6413.6   78.55  6416.1   78.54
  6453.6    78.4  6466.1   78.53  6503.6   78.91  6513.6   79.54  6516.1   79.56
  6543.6   79.83  6573.6   80.85  6593.6   82.18  6596.1   82.27  6623.9   83.21
  6673.6    84.9  6693.6   86.37  6701.7   86.63
BR D #Mann= 3
 2786.80   0.135  4976.5    0.05  5023.5   0.135
BR D Banks=4976.50,5023.50

Type RM Length L Ch R = 1 ,149160.8,644.2,644.2,644.2
BEGIN DESCRIPTION:
Downstream Section of Bridge/Culvert/Weir
END DESCRIPTION:
#Sta/Elev= 30
  2786.8    89.5  3711.1   80.02  4391.2   78.79  4431.2   75.84  4560.4   76.83
  4590.4   76.04  4600.4   76.75  4767.6   76.09  4937.6   74.13  4976.5      73
    4980   67.91    5020   67.91  5023.5      73  5067.6   74.06    5108   72.87
    5198   72.66    5228   74.27    5298   74.95    5318   73.85    5408   74.99
  5663.6   74.28  5713.6   73.47  5793.6    74.2  5853.6   77.14  5943.6    74.9
  6083.6   77.57  6453.6    78.4  6543.6   79.83  6673.6    84.9  6701.7   86.63
#Mann= 3 , 1 , 0
 2786.80   0.135       0  4976.5    0.05       0  5023.5   0.135       0
#XS Ineff= 2 , 0
       0 4969.83   78.01 5030.17       0   76.83
Bank Sta=4976.50,5023.50
Exp/Cntr=0.5,0.3

Type RM Length L Ch R = 1 ,148516.6,499.3,499.3,499.3
BEGIN DESCRIPTION:
Town Creek 295.0
END DESCRIPTION:
#Sta/Elev= 30
  2779.4   96.68  2839.4   91.35  2959.4   85.96  3169.4   82.11  3239.4    83.2
  3469.4   76.88  3549.4   79.53  3629.4   78.52  3709.4   80.29  3989.4   77.65
  4339.4   77.85  4399.4    73.8  4439.4   73.22  4579.4   73.94  4639.4   78.45
  4789.4   78.45  4899.4   72.19 4978.44   70.89 4979.49   67.89 5020.58   67.89
 5021.63   70.89    5060    74.8    5160   73.29    5260   76.83    5570   74.44
    5840   76.03    5970   74.04    6010   78.49    6110   94.33  6225.4   95.85
#Mann= 3 , 1 , 0
 2779.40   0.142       0 4978.44    0.05       0 5021.63   0.142       0
Bank Sta=4978.44,5021.63
Exp/Cntr=0.3,0.1

Type RM Length L Ch R = 1 ,148017.3,499.8,499.8,499.8
BEGIN DESCRIPTION:
Town Creek 294.0
END DESCRIPTION:
#Sta/Elev= 30
  4367.7   81.38  4488.5   79.61  4518.5   80.16  4568.5   77.44  4618.5   77.69
  4718.5   74.63  4758.5   75.67  4788.5   75.65  4798.5   76.48  4818.5   75.93
  4848.5   76.44  4918.5   72.92  4958.5   72.65 4978.37   70.88 4979.42   67.88
 5020.51   67.88 5021.56   70.88    5150   74.42    5170   75.55    5220   73.66
    5640   74.52    5670   73.39    5740   73.94    5810   73.05    5860   73.97
    5920   78.01    6000   87.72    6010   87.62    6090   91.84  6122.2   92.88
#Mann= 3 , 1 , 0
 4367.70   0.142       0 4978.37    0.05       0 5021.56   0.142       0
Bank Sta=4978.37,5021.56
Exp/Cntr=0.3,0.1

Type RM Length L Ch R = 1 ,147517.5,499.4,499.4,499.4
BEGIN DESCRIPTION:
Town Creek 293.0
END DESCRIPTION:
#Sta/Elev= 30
  4079.5    81.5  4319.5   79.27  4429.5   79.29  4499.5    77.8  4579.5    74.4
  4669.5   75.26  4699.5   73.77  4969.5   74.31 4978.37   70.88 4979.42   67.88
 5020.51   67.88 5021.56   70.88    5060   73.96    5110   72.54    5170    72.1
    5210   72.46    5230   73.27    5270   72.52    5290    73.2    5330   73.24
    5380   72.36    5560   72.57    5640   75.28    5740   82.39    5760   82.73
    5810   86.91    5850   88.02    5900   90.92    5910    90.3  5970.3   91.01
#Mann= 3 , 1 , 0
 4079.50   0.142       0 4978.37    0.05       0 5021.56   0.142       0
Bank Sta=4978.37,5021.56
Exp/Cntr=0.3,0.1

Type RM Length L Ch R = 1 ,147018.1,688.7,688.7,688.7
BEGIN DESCRIPTION:
Town Creek 292.0
END DESCRIPTION:
#Sta/Elev= 26
  4316.2    81.6    4320   81.44  4396.2   78.15  4436.2   77.93  4476.2   75.43
  4566.2   73.51  4806.2   75.63  4866.2   75.99 4978.44   70.87 4979.49   67.87
 5020.58   67.87 5021.63   70.87    5120   73.85    5140   74.77    5220   74.76
    5310   73.96    5400   71.91    5600   73.59    5610    73.4    5660   74.71
    5810   94.33    5820   95.29    5860    96.1    5880   97.79    5930   96.97
  6040.9   97.94
#Mann= 4 , 1 , 0
 4316.20    0.19       0    4320   0.142       0 4978.44    0.05       0
 5021.63   0.142       0
Bank Sta=4978.44,5021.63
Exp/Cntr=0.3,0.1

Type RM Length L Ch R = 1 ,146329.4,1076.7,1076.7,1076.7
BEGIN DESCRIPTION:
Town Creek 290.0
END DESCRIPTION:
#Sta/Elev= 29
  4154.9   81.29  4314.9   75.31  4424.9   75.85  4514.9      73  4604.9   72.94
  4664.9   72.24  4684.9   72.57  4705.8   72.49  4975.8   72.83 4978.37   70.86
 4979.42   67.86 5020.51   67.86 5021.56   70.86  5045.8    72.7  5075.8   74.33
  5225.8    74.1  5265.8   74.69  5345.8   71.66  5485.8   73.12  5505.8   73.76
  5535.8   73.16  5625.8   73.94  5635.8   74.32  5665.8   77.39  5675.8   78.91
  5685.8   80.99  5745.8   89.24  5785.8   92.36  5911.3   93.11
#Mann= 3 , 1 , 0
 4154.90   0.142       0 4978.37    0.05       0 5021.56   0.142       0
Bank Sta=4978.37,5021.56
Exp/Cntr=0.3,0.1

Type RM Length L Ch R = 1 ,145252.7,580.7,580.7,580.7
BEGIN DESCRIPTION:
Town Creek 289.0
END DESCRIPTION:
#Sta/Elev= 30
  4480.6   78.28    4485   78.24  4550.6   77.61  4580.6   76.64  4650.6      76
  4660.6   76.27  4720.6   73.82  4780.6    73.5  4800.6   72.64  4970.6   72.68
 4977.53   70.83 4978.58   67.83 5021.49   67.83 5022.54   70.83  5241.9   72.88
  5261.9   72.17  5401.9    72.4  5501.9   74.91  5661.9   73.99  5771.9   75.15
  5811.9   74.47  5861.9   74.67  5971.9    78.2  6071.9   76.56  6221.9   78.32
  6291.9   76.98  6391.9   80.41  6421.9   80.29  6551.9   90.94  6697.6   92.99
#Mann= 4 , 1 , 0
 4480.60    0.19       0    4485   0.142       0 4977.53    0.05       0
 5022.54   0.142       0
Bank Sta=4977.53,5022.54
Exp/Cntr=0.3,0.1

Type RM Length L Ch R = 1 ,144672.0,705.8,705.8,705.8
BEGIN DESCRIPTION:
Town Creek 288.0
END DESCRIPTION:
#Sta/Elev= 30
  3367.9   83.88  3917.9   79.07  4167.9   79.02  4227.9   77.17  4287.9   73.08
  4317.9   72.63  4347.9    73.8  4557.9   72.41  4677.9   73.65  4707.9   72.85
  4747.9   74.04  4847.9   74.69  4887.9   73.46  4927.9   73.39 4977.53    70.6
 4978.58    67.6 5021.49    67.6 5022.54    70.6    5037   71.75    5367   73.31
    5427   71.92    5767   73.12    5787   72.64    5897   77.57    6047   75.24
    6167   76.71    6437   83.81    6597   91.91    6647   91.06  6713.8   92.07
#Mann= 3 , 1 , 0
 3367.90   0.142       0 4977.53    0.05       0 5022.54   0.142       0
Bank Sta=4977.53,5022.54
Exp/Cntr=0.3,0.1

Type RM Length L Ch R = 1 ,143966.2,452.6,452.6,452.6
BEGIN DESCRIPTION:
Town Creek 287.0
END DESCRIPTION:
#Sta/Elev= 30
  3524.3   84.38  3894.3   80.56  4204.3   78.63  4264.3   74.03  4374.3    72.5
  4454.3    73.3  4894.3   72.89 4977.53   70.44 4978.58   67.44 5021.49   67.44
 5022.54   70.44  5024.3   72.12  5080.2   72.96  5090.2   72.36  5110.2   73.17
  5140.2   72.71  5160.2   71.65  5370.2   72.09  5420.2   74.49  5580.2   74.33
  5620.2   72.42  5818.8    77.5  5988.8   78.77  6098.8   78.72  6398.8   76.61
  6468.8   78.57  6658.8   87.13  6838.8   89.07  7158.8    98.6  7245.4   99.85
#Mann= 3 , 1 , 0
 3524.30   0.142       0 4977.53    0.05       0 5022.54   0.142       0
Bank Sta=4977.53,5022.54
Exp/Cntr=0.3,0.1

Type RM Length L Ch R = 1 ,143513.6,499.3,499.3,499.3
BEGIN DESCRIPTION:
Town Creek 286.0
END DESCRIPTION:
#Sta/Elev= 30
  3504.3   86.72  3744.3   81.93  3934.3   79.44  4134.3   78.95  4214.3    72.4
  4234.3   72.17  4284.3   72.99  4364.3   71.63  4674.3   71.45  4904.3   72.77
  4964.3      72 4977.53   70.35 4978.58   67.35 5021.49   67.35 5022.54   70.35
    5040   72.63    5110   71.22    5180   72.82    5200   71.82    5460   71.75
    5490   73.36    5650   73.59    5670   72.75    5900   72.09    5950   75.66
    6020   77.15    6070   75.33    6190   77.19    6240   76.69  6335.2   80.03
#Mann= 3 , 1 , 0
 3504.30   0.142       0 4977.53    0.05       0 5022.54   0.142       0
Bank Sta=4977.53,5022.54
Exp/Cntr=0.3,0.1

Type RM Length L Ch R = 1 ,143014.3,500.5,500.5,500.5
BEGIN DESCRIPTION:
Town Creek 285.0
END DESCRIPTION:
#Sta/Elev= 30
  3774.9   83.62  3844.9   81.65  3934.9   80.68  4114.9   79.94  4194.9   73.46
  4234.9   72.97  4434.9   73.27  4474.9   72.44 4977.46   70.24 4978.51   67.24
 5021.42   67.24 5022.47   70.24    5040   72.09    5420    71.3    5500   71.48
    5530    72.3    5690   70.41    5840   72.78    5870   74.41    5940   74.28
    5970   72.08    6160   70.84    6180   72.15    6220   77.69  6324.2   79.79
  7084.2   76.69  7134.2   79.04  7224.2   79.23  7334.2   82.18  7440.2   88.34
#Mann= 3 , 1 , 0
 3774.90   0.142       0 4977.46    0.05       0 5022.47   0.142       0
Bank Sta=4977.46,5022.47
Exp/Cntr=0.3,0.1

Type RM Length L Ch R = 1 ,142513.8,500.9,500.9,500.9
BEGIN DESCRIPTION:
Town Creek 284.0
END DESCRIPTION:
#Sta/Elev= 27
  3695.9   82.27  3745.9   81.52  3755.9   81.79  3935.9   78.65  3975.9   75.72
  4005.9    74.3  4125.9   75.55  4235.9   72.88  4245.9   72.94  4275.9   72.02
  4345.9    73.5  4435.9   71.98  4505.9   73.61  4575.9   73.17  4615.9    71.6
  4745.9    70.7  4945.9   71.01 4977.53   69.66 4978.58   66.66 5021.49   66.66
 5022.54   69.66    5200    69.6    5270   70.56    5750   71.58    5910   76.86
    6280   77.72    6490   78.24
#Mann= 3 , 1 , 0
 3695.90   0.142       0 4977.53    0.05       0 5022.54   0.142       0
Bank Sta=4977.53,5022.54
Exp/Cntr=0.3,0.1

Type RM Length L Ch R = 1 ,142012.9,500.4,500.4,500.4
BEGIN DESCRIPTION:
Town Creek 283.0
END DESCRIPTION:
#Sta/Elev= 20
  3834.1   83.09  4494.1   74.19  4524.1   73.04  4554.1   73.13  4594.1   71.84
  4804.1   69.72  4884.1   70.76 4977.46   69.49 4978.51   66.49 5021.42   66.49
 5022.47   69.49    5040   70.47    5070   69.83    5170      75    5400   73.29
    5540   75.15    5640   73.85    5950   76.86    5970   76.53    6030   77.12
#Mann= 3 , 1 , 0
 3834.10   0.142       0 4977.46    0.05       0 5022.47   0.142       0
Bank Sta=4977.46,5022.47
Exp/Cntr=0.3,0.1

Type RM Length L Ch R = 1 ,141512.5,551.7,551.7,551.7
BEGIN DESCRIPTION:
Town Creek 282.0
END DESCRIPTION:
#Sta/Elev= 21
  3626.1   85.68  3636.1   85.85  4196.1   78.58  4226.1   75.39  4286.1   74.06
  4386.1   73.83  4566.1   75.29  4666.1   70.63  4976.1    70.6 4977.46   69.06
 4978.51   66.06 5021.42   66.06 5022.47   69.06    5040    70.3    5110   69.82
    5550   70.41    5620    74.4    6050   76.66    6160   77.23    6330   77.57
    6380   77.67
#Mann= 4 , 1 , 0
 3626.10   0.135       0 4977.46    0.05       0 5022.47   0.135       0
    6330    0.18       0
Bank Sta=4977.46,5022.47
Exp/Cntr=0.3,0.1

Type RM Length L Ch R = 1 ,140960.8,446.9,446.9,446.9
BEGIN DESCRIPTION:
Town Creek 281.0
END DESCRIPTION:
#Sta/Elev= 30
  3641.4   90.25  3661.4   90.15  3711.4   87.29  3731.4    87.7  3801.4   84.95
  3951.4   82.81  3981.4   81.48  4091.4   72.69  4121.4    72.5  4201.4   74.63
  4771.4   69.96  4931.4   70.44  4941.4   69.11 4977.53   68.94 4978.58   65.94
 5021.49   65.94 5022.54   68.94  5319.2   70.29  5349.2   69.18  5379.2   70.19
  5609.2   69.57  5719.2   72.83    5852   74.35    5932   73.42    6042    69.8
    6112   71.31    6162   74.52    6332   75.02    6412   81.73  6501.2   85.86
#Mann= 3 , 1 , 0
 3641.40   0.135       0 4977.53    0.05       0 5022.54   0.135       0
Bank Sta=4977.53,5022.54
Exp/Cntr=0.3,0.1

Type RM Length L Ch R = 1 ,140513.9,498.8,498.8,498.8
BEGIN DESCRIPTION:
Town Creek 280.0
END DESCRIPTION:
#Sta/Elev= 30
  3804.5   92.13  4024.5   83.66  4064.5   83.73  4144.5   78.88  4184.5   78.15
  4254.5   73.34  4324.5   71.79  4454.5   73.07  4514.5   71.92  4564.5   70.31
  4704.5   73.53  4814.5    73.6  4914.5   71.35  4944.5    69.8 4977.46   68.87
 4978.51   65.87 5021.42   65.87 5022.47   68.87    5230   70.19    5470   69.68
    5490   70.46    5730   71.26    5750   70.88    5860   72.18    5970   71.75
    5990   72.59    6080   73.46    6190   79.82    6220   82.35  6358.1   87.01
#Mann= 3 , 1 , 0
 3804.50   0.135       0 4977.46    0.05       0 5022.47   0.135       0
Bank Sta=4977.46,5022.47
Exp/Cntr=0.3,0.1

Type RM Length L Ch R = 1 ,140015.1,499.4,499.4,499.4
BEGIN DESCRIPTION:
Town Creek 279.0
END DESCRIPTION:
#Sta/Elev= 28
  3560.8   95.58  3580.8   95.52  3650.8   91.26  3720.8   81.92  3820.8   76.87
  3950.8   74.55  4090.8   75.99  4170.8   73.16  4200.8   72.92  4230.8    71.5
  4350.8   70.24  4390.8   71.12  4640.8    70.4  4970.8   70.54 4977.46   68.85
 4978.51   65.85 5021.42   65.85 5022.47   68.85    5520   72.61  5614.6   73.58
  5674.6   74.94  5804.6   74.86  5844.6   75.85  5904.6   76.83  5994.6   82.48
  6034.6   83.93  6214.6   86.09  6466.3   90.49
#Mann= 3 , 1 , 0
 3560.80   0.135       0 4977.46    0.05       0 5022.47   0.135       0
Bank Sta=4977.46,5022.47
Exp/Cntr=0.3,0.1

Type RM Length L Ch R = 1 ,139515.7,499,499,499
BEGIN DESCRIPTION:
Town Creek 278.0
END DESCRIPTION:
#Sta/Elev= 28
  3542.6    99.6  3572.6   98.13  3592.6   98.06  3902.6   77.34  3992.6   74.05
  4292.6    70.4  4362.6   70.11  4712.6   70.22  4882.6   70.13  4892.6   69.66
 4977.53   68.82 4978.58   65.82 5021.49   65.82 5022.54   68.82    5150    70.3
    5200   69.74    5280   70.15    5360   69.64    5530   72.61    5720   74.49
    5740   74.03    5810   74.77    5830   76.55    5880   79.01    5910   80.37
    6080   82.59    6360   89.22  6458.6   89.37
#Mann= 3 , 1 , 0
 3542.60   0.135       0 4977.53    0.05       0 5022.54   0.135       0
Bank Sta=4977.53,5022.54
Exp/Cntr=0.3,0.1

Type RM Length L Ch R = 1 ,139016.7,499.4,499.4,499.4
BEGIN DESCRIPTION:
Town Creek 277.0
END DESCRIPTION:
#Sta/Elev= 27
  3533.7   93.55  3623.7    88.7  3643.7   85.94  3653.7   85.05  3673.7   84.43
  3713.7    80.6  3793.7   76.89  3933.7      75  4103.7   73.65  4153.7   70.91
  4273.7   69.96  4393.7   70.08  4583.7   71.86  4713.7   70.23  4723.7   70.55
  4943.7   70.25 4977.53   68.78 4978.58   65.78 5021.42   65.78 5022.47   68.78
    5030   70.24    5240   70.08    5300   74.42    5630   74.63    5660   75.47
    6290    82.2  6574.2   85.01
#Mann= 3 , 1 , 0
 3533.70   0.135       0 4977.53    0.05       0 5022.47   0.135       0
Bank Sta=4977.53,5022.47
Exp/Cntr=0.3,0.1

Type RM Length L Ch R = 1 ,138517.3,500.6,500.6,500.6
BEGIN DESCRIPTION:
Town Creek 276.0
END DESCRIPTION:
#Sta/Elev= 26
  3695.9   90.24  3835.9   75.82  3865.9   73.95  4025.9   70.89  4055.9   71.53
  4245.9   71.66  4355.9   69.98  4395.9   70.51  4415.9   69.78  4605.9   71.02
  4645.9   69.43  4735.9   70.32  4865.9   70.48  4905.9   71.61  4975.9   70.17
 4977.46   68.74 4978.51   65.74 5021.42   65.74 5022.47   68.74    5330   70.02
    5360   70.75    5600   70.48    5890   78.56    6330   78.46    6350    80.9
  6462.4   82.17
#Mann= 3 , 1 , 0
 3695.90   0.135       0 4977.46    0.05       0 5022.47   0.135       0
Bank Sta=4977.46,5022.47
Exp/Cntr=0.3,0.1

Type RM Length L Ch R = 1 ,138016.7,499.4,499.4,499.4
BEGIN DESCRIPTION:
Town Creek 275.0
END DESCRIPTION:
#Sta/Elev= 30
  3600.2   91.27  3640.2   87.87  3780.2   80.32  3870.2   77.65  3890.2   76.48
  4020.2   73.68  4050.2   72.06  4220.2   69.41  4370.2   71.42  4660.2   69.89
  4740.2   70.19  4770.2   68.86  4850.2   69.98  4860.2   69.71 4977.46    68.7
 4978.51    65.7 5021.42    65.7 5022.47    68.7    5100   70.41    5350   70.08
    5390   69.02    5450   69.78    5750   69.93    5770    70.9    5790   72.95
    6070   78.74    6290   78.09    6350   78.28    6390   80.88  6434.6   81.12
#Mann= 3 , 1 , 0
 3600.20   0.135       0 4977.46    0.05       0 5022.47   0.135       0
Bank Sta=4977.46,5022.47
Exp/Cntr=0.3,0.1

Type RM Length L Ch R = 1 ,137517.3,499.2,499.2,499.2
BEGIN DESCRIPTION:
Town Creek 274.0
END DESCRIPTION:
#Sta/Elev= 29
  3390.8   89.11  3700.8   78.92  3720.8   77.55  3740.8   77.26  3810.8   72.06
  3830.8   72.29  3860.8   70.03  3980.8   70.01  4000.8   69.61  4090.8   70.35
  4440.8   69.35  4540.8   70.12  4580.8   69.48 4977.46   68.66 4978.51   65.66
 5021.42   65.66 5022.47   68.66    5060   69.97    5090   71.18    5270   69.52
    5510   69.14    5530   68.65    5540   70.09    5600   72.04    5750   73.09
    6060   70.72    6070   72.36    6250    75.5  6458.6   80.52
#Mann= 3 , 1 , 0
 3390.80   0.135       0 4977.46    0.05       0 5022.47   0.135       0
Bank Sta=4977.46,5022.47
Exp/Cntr=0.3,0.1

Type RM Length L Ch R = 1 ,137018.1,499.8,499.8,499.8
BEGIN DESCRIPTION:
Town Creek 273.0
END DESCRIPTION:
#Sta/Elev= 27
  3501.3   88.45  3531.3   87.85  3731.3   81.08  3901.3   76.62  3991.3   69.94
  4191.3    70.2  4211.3   70.76  4851.3   68.31  4881.3   69.19 4977.53   68.62
 4978.58   65.62 5021.49   65.62 5022.54   68.62    5180   68.97    5310   69.47
    5330   68.95    5370   68.85    5530   68.96    5570   71.56    5640    73.2
    5750   71.96    5780   72.44    6030   72.29    6050    72.3    6170   75.21
    6390   83.37  6447.7   84.08
#Mann= 4 , 1 , 0
 3501.30   0.135       0 4977.53    0.05       0 5022.54   0.135       0
    5640    0.18       0
Bank Sta=4977.53,5022.54
Exp/Cntr=0.3,0.1

Type RM Length L Ch R = 1 ,136518.3,711.1,711.1,711.1
BEGIN DESCRIPTION:
Town Creek 272.0
END DESCRIPTION:
#Sta/Elev= 30
  3682.2   78.65  3872.2   74.51  3972.2    69.8  4122.2   68.42  4202.2   69.75
  4322.2    68.3  4382.2   69.25  4572.2    68.4 4977.46   68.58 4978.51   65.58
 5021.42   65.58 5022.47   68.58    5450   69.54    5490   68.24    5600   69.16
    5680   70.76    5880   72.17    5900   73.07    5950   72.95    6040   75.46
    6100   78.53    6120   78.87    6130   80.49    6140   83.53    6150   87.68
    6160   88.97    6170   87.69    6180   85.02    6190   83.94    6242   83.93
#Mann= 3 , 1 , 0
 3682.20   0.135       0 4977.46    0.05       0 5022.47   0.135       0
Bank Sta=4977.46,5022.47
Exp/Cntr=0.3,0.1

Type RM Length L Ch R = 1 ,135807.2,534.3,534.3,534.3
BEGIN DESCRIPTION:
Town Creek 271.0
END DESCRIPTION:
#Sta/Elev= 30
  3117.3   86.79  3267.3   84.58  3357.3   80.23  3407.3   82.52  3477.3   78.46
  3487.3   79.34  3767.3   73.04  3937.3    73.9  4027.3    69.2  4037.3    67.6
  4147.3   67.47  4177.3   68.48 4976.76    67.4 4977.81    64.4 5022.12    64.4
 5023.17    67.4  5278.1   70.71  5418.1   69.73  5738.1   73.54  5878.1   78.59
  5918.1   88.45  5928.1   88.18  5948.1   84.03  6138.1    83.3  6158.1      87
  6168.1   91.26  6208.1   92.16  6218.1   94.59  6248.1   96.65  6293.7   95.94
#Mann= 3 , 1 , 0
 3117.30   0.135       0 4976.76    0.05       0 5023.17   0.135       0
Bank Sta=4976.76,5023.17
Exp/Cntr=0.3,0.1

Type RM Length L Ch R = 1 ,135272.9,755.9,755.9,755.9
BEGIN DESCRIPTION:
Town Creek 269.0
END DESCRIPTION:
#Sta/Elev= 30
  3706.2   84.95  3766.2   84.85  3886.2   74.91  4326.2   71.48  4396.2   68.31
  4446.2   69.38  4626.2   65.92  4696.2   66.88  4756.2   66.14 4976.83   65.84
 4977.88   62.84 5022.19   62.84 5023.24   65.84  5296.2   67.39  5316.2   66.87
  5384.4      69  5494.4    67.3  5744.4   72.78  5974.4   73.18  6054.4   75.18
  6144.4   73.06  6184.4   73.36  6254.4   77.05  6284.4   80.58  6304.4   87.08
  6344.4   93.33  6354.4   95.53  6374.4   98.08  6424.4   99.73  6503.4  101.17
#Mann= 3 , 1 , 0
 3706.20   0.128       0 4976.83    0.05       0 5023.24   0.128       0
Bank Sta=4976.83,5023.24
Exp/Cntr=0.3,0.1

Type RM Length L Ch R = 1 ,134517.0,500,500,500
BEGIN DESCRIPTION:
Town Creek 268.0
END DESCRIPTION:
#Sta/Elev= 30
  3729.2   89.83  3829.2   87.91  3889.2   85.53  3909.2   83.62  3939.2    78.6
  3989.2   74.51  4029.2   72.54  4529.2   66.42  4639.2   68.83  4939.2   65.71
  4969.2   66.55 4976.76    65.8 4977.81    62.8 5022.12    62.8 5023.17    65.8
    5060    66.9    5180   65.68    5760   67.71    5860   71.41    6190   73.14
    6310   72.02    6330   73.34    6360   72.91    6440   74.92    6580    72.3
    6680   77.28    6830   90.74    6870   96.34    6940  102.27  6952.2  104.17
#Mann= 3 , 1 , 0
 3729.20   0.128       0 4976.76    0.05       0 5023.17   0.128       0
Bank Sta=4976.76,5023.17
Exp/Cntr=0.3,0.1

Type RM Length L Ch R = 1 ,134017.0,500,500,500
BEGIN DESCRIPTION:
Town Creek 267.0
END DESCRIPTION:
#Sta/Elev= 30
  3580.3   87.56  3620.3    86.4  3650.3   84.33  3690.3   83.45  3810.3   73.69
  3860.3   72.22  4450.3   72.33  4490.3   70.86  4610.3   69.93  4680.3   66.55
  4820.3   65.51  4860.3   66.49 4976.83   65.78 4977.88   62.78 5022.19   62.78
 5023.24   65.78    5190    65.7    5310    66.9    5330   66.43    5440   65.52
    5500   67.28    5770   67.57    6140   70.38    6170   69.42    6210   69.87
    6240   71.59    6350   85.88    6380   87.62    6450   89.02    6623   93.68
#Mann= 3 , 1 , 0
 3580.30   0.128       0 4976.83    0.05       0 5023.24   0.128       0
Bank Sta=4976.83,5023.24
Exp/Cntr=0.3,0.1

Type RM Length L Ch R = 1 ,133517.0,499.1,499.1,499.1
BEGIN DESCRIPTION:
Town Creek 266.0
END DESCRIPTION:
#Sta/Elev= 30
  3587.6   92.95  3677.6   87.77  3787.6   75.63  4137.6   71.13  4397.6   71.93
  4417.6   70.74  4447.6   71.11  4627.6   68.15  4707.6   69.24  4747.6   70.92
  4907.6   65.82 4976.83   65.07 4977.88   62.07 5022.19   62.07 5023.24   65.07
    5240   66.78    5340    65.3    5440   66.47    5940   67.38    6030   66.39
    6170   67.46    6250   74.71  6380.3   72.67  6400.3   71.35  6520.3   73.11
  6610.3   79.16  6680.3   86.68  6720.3   87.53  6760.3   91.34  6779.7   91.31
#Mann= 3 , 1 , 0
 3587.60   0.128       0 4976.83    0.05       0 5023.24   0.128       0
Bank Sta=4976.83,5023.24
Exp/Cntr=0.3,0.1

Type RM Length L Ch R = 1 ,133017.9,499.2,499.2,499.2
BEGIN DESCRIPTION:
Town Creek 265.0
END DESCRIPTION:
#Sta/Elev= 29
  3534.1   81.35  3554.1   79.62  3654.1   75.48  3934.1   71.73  4114.1   72.78
  4244.1   67.87  4344.1    70.6  4384.1   69.48  4444.1   66.27  4524.1   65.55
  4534.1    65.9  4754.1   67.28  4834.1   65.21 4976.83   64.08 4977.88   61.08
 5022.19   61.08 5023.24   64.08    5140   64.79    5160   65.65    5210   64.42
    5230   64.85    5260    64.2    5410    67.7    5490   66.14    5700   68.03
    5930   76.84    6000   78.14    6040   78.53  6115.1   82.75
#Mann= 3 , 1 , 0
 3534.10   0.128       0 4976.83    0.05       0 5023.24   0.128       0
Bank Sta=4976.83,5023.24
Exp/Cntr=0.3,0.1

Type RM Length L Ch R = 1 ,132518.7,499.6,499.6,499.6
BEGIN DESCRIPTION:
Town Creek 264.0
END DESCRIPTION:
#Sta/Elev= 24
  3222.8   90.59  3292.8   89.14  3572.8   70.49  3602.8   69.99  3642.8   68.01
  3672.8   68.78  3782.8   66.46  3882.8   66.45  3962.8   65.45  4462.8   68.19
  4552.8    64.8  4732.8   66.08  4842.8   65.02  4922.8   65.78  4942.8   65.32
  4952.8   65.58 4976.83   63.99 4977.88   60.99 5022.12   60.99 5023.17   63.99
    5200   64.62    5490    66.4    5760   80.54  5776.7   81.01
#Mann= 3 , 1 , 0
 3222.80   0.128       0 4976.83    0.05       0 5023.17   0.128       0
Bank Sta=4976.83,5023.17
Exp/Cntr=0.3,0.1

Type RM Length L Ch R = 1 ,132019.1,499.5,499.5,499.5
BEGIN DESCRIPTION:
Town Creek 263.0
END DESCRIPTION:
#Sta/Elev= 30
  3235.5   101.7  3375.5   95.57  3455.5   89.58  3495.5   83.16  3525.5   80.52
  3765.5   72.76  3815.5    69.3  3845.5    65.6  4065.5   65.96  4135.5   68.54
  4205.5   67.58  4255.5   65.69  4345.5    64.9  4465.5   65.68  4695.5   64.64
  4805.5   66.56  4865.5   64.53  4955.5      65 4976.83   63.89 4977.88   60.89
 5022.19   60.89 5023.24   63.89    5070   64.94    5420   67.25    5580   65.64
    5740   70.58    5970   74.57    6080   80.81    6170   88.74  6279.9   91.51
#Mann= 3 , 1 , 0
 3235.50   0.128       0 4976.83    0.05       0 5023.24   0.128       0
Bank Sta=4976.83,5023.24
Exp/Cntr=0.3,0.1

Type RM Length L Ch R = 1 ,131519.6,500.8,500.8,500.8
BEGIN DESCRIPTION:
Town Creek 262.0
END DESCRIPTION:
#Sta/Elev= 30
    3430  100.55    3530   96.89    3610   88.47    3620   86.83    3720   79.25
    3880   74.49    4070   71.42    4110   66.59    4170   64.81    4370   67.45
    4440   65.69    4970   64.83 4976.83   63.78 4977.88   60.78 5022.19   60.78
 5023.24   63.78    5030   64.71    5160   65.37    5240   64.07    5470   64.76
    5720   66.73    5770   65.83    5850   67.76    5910   70.47    6060   72.03
    6080   71.01    6220   73.19    6270   76.05    6390   85.13  6408.6   85.68
#Mann= 3 , 1 , 0
 3430.00   0.128       0 4976.83    0.05       0 5023.24   0.128       0
Bank Sta=4976.83,5023.24
Exp/Cntr=0.3,0.1

Type RM Length L Ch R = 1 ,131018.8,499.5,499.5,499.5
BEGIN DESCRIPTION:
Town Creek 261.0
END DESCRIPTION:
#Sta/Elev= 30
  3147.5  102.05  3317.5   96.11  3357.5   90.85  3457.5   87.34  3547.5   79.02
  3697.5   73.66  3807.5   72.01  3897.5   68.12  3997.5   66.54  4177.5   67.91
  4237.5   65.07  4417.5   65.52  4447.5   66.74  4487.5    70.6  4547.5   67.98
  4627.5   67.87  4737.5   64.98 4976.76   63.68 4977.81   60.68 5022.12   60.68
 5023.17   63.68    5150      65    5550   64.81    5880   66.95    5990   75.22
    6010   79.47    6070   75.33    6120   75.19    6200   77.74  6369.6   76.95
#Mann= 3 , 1 , 0
 3147.50   0.128       0 4976.76    0.05       0 5023.17   0.128       0
Bank Sta=4976.76,5023.17
Exp/Cntr=0.3,0.1

Type RM Length L Ch R = 1 ,130519.3,999.1,999.1,999.1
BEGIN DESCRIPTION:
Town Creek 260.0
END DESCRIPTION:
#Sta/Elev= 30
  2735.9   102.1  2775.9   101.8  2925.9   95.56  2955.9   93.03  3005.9   90.59
  3025.9   88.15  3095.9   85.55  3115.9   83.08  3195.9   78.87  3265.9   77.02
  3295.9   77.32  3505.9   70.93  3535.9   69.09  3745.9   70.65  3935.9   67.78
  4185.9   70.51  4725.9   67.86  4805.9   64.65 4976.76   63.57 4977.81   60.57
 5022.12   60.57 5023.17   63.57    5280   64.99    5380   63.56    5590   64.23
    5750   66.15    5840   65.41    5850   65.78    5960   82.91  6150.7   85.31
#Mann= 3 , 1 , 0
 2735.90   0.128       0 4976.76    0.05       0 5023.17   0.128       0
Bank Sta=4976.76,5023.17
Exp/Cntr=0.3,0.1

Type RM Length L Ch R = 1 ,129520.2,843.2,843.2,843.2
BEGIN DESCRIPTION:
Town Creek 259.0
END DESCRIPTION:
#Sta/Elev= 30
  3578.3   82.95  3778.3   76.61  3858.3   75.66  3878.3   74.19  3938.3      72
  3958.3   70.76  4018.3   68.93  4028.3   68.22  4348.3   70.61  4458.3   69.03
  4538.3   70.57  4778.3   67.02  4828.3   64.19  4968.3   64.55 4976.76   63.37
 4977.81   60.37 5022.12   60.37 5023.17   63.37    5030   64.08    5730   63.86
    5750    63.5    5820   64.89    6000    64.3    6040   63.44    6060   65.36
    6120   63.89    6130    64.2    6150    63.8    6190   67.38  6620.9   73.58
#Mann= 3 , 1 , 0
 3578.30   0.128       0 4976.76    0.05       0 5023.17   0.128       0
Bank Sta=4976.76,5023.17
Exp/Cntr=0.3,0.1

Type RM Length L Ch R = 1 ,128677.0,776,776,776
BEGIN DESCRIPTION:
Town Creek 257.0
END DESCRIPTION:
#Sta/Elev= 30
  3185.6   95.92  3345.6   86.85  3355.6   87.04  3375.6   84.89  3825.6   75.73
  4085.6   71.54  4185.6   68.26  4545.4   68.56  4825.4   65.78  4855.4   64.66
 4976.76   62.89 4977.81   59.89 5022.12   59.89 5023.17   62.89  5105.4   65.54
  5175.4    63.2  5552.4    63.6  5582.4   64.94  5632.4   65.56  5652.4   64.65
  5752.4   63.53  5772.4   64.67  5802.4   63.89  5882.4   63.92  5962.4    69.2
  6042.4   69.24  6472.4   73.25  6522.4   76.93  6572.4   78.06  6602.5   79.39
#Mann= 3 , 1 , 0
 3185.60   0.128       0 4976.76    0.05       0 5023.17   0.128       0
Bank Sta=4976.76,5023.17
Exp/Cntr=0.3,0.1

Type RM Length L Ch R = 1 ,127901.0,1383.1,1383.1,1383.1
BEGIN DESCRIPTION:
Town Creek 255.0
END DESCRIPTION:
#Sta/Elev= 30
  2773.9   96.48  2843.9   96.37  2933.9   92.27  3063.9   83.21  3383.9   76.32
  3563.9   75.68  4123.9   68.16  4323.9   70.27  4653.9   67.68  4831.2   63.47
  4971.2   62.92 4976.76   62.01 4977.81   59.01 5022.12   59.01 5023.17   62.01
  5041.2   64.53  5101.2   63.83  5121.2    62.8  5251.2   62.51  5281.2    63.6
  5321.2    62.4  5411.2   62.17  5491.2   63.34  5521.2   62.69  5841.2   64.39
  5891.2   65.66  5921.2   69.21  5971.2   71.01  6031.2   70.92  6323.1    76.9
#Mann= 3 , 1 , 0
 2773.90   0.128       0 4976.76    0.05       0 5023.17   0.128       0
Bank Sta=4976.76,5023.17
Exp/Cntr=0.3,0.1

Type RM Length L Ch R = 1 ,126517.9,501.3,501.3,501.3
BEGIN DESCRIPTION:
Town Creek 253.0
END DESCRIPTION:
#Sta/Elev= 30
  1285.3   82.51  1875.3    75.5  2105.3   76.18  2115.3   74.31  2135.3   75.79
  2865.3    75.2  3305.3   68.61  3515.3   68.39  3535.3   69.39  3575.3   67.57
  3855.3   66.44  3895.3   64.79  3955.3   66.92  4175.3   63.36  4255.3   64.49
  4345.3   68.62  4405.3   62.92  4445.3   67.37  4515.3   63.53  4625.3      67
  4785.3   67.76  4855.3   63.07 4975.57   61.05 4976.62   58.05 5023.45   58.05
  5024.5   61.05    5560   61.85    5640   69.54    5840   96.96  5887.5  101.68
#Mann= 3 , 1 , 0
 1285.30    0.15       0 4975.57    0.05       0  5024.5    0.15       0
Bank Sta=4975.57,5024.50
Exp/Cntr=0.3,0.1

Type RM Length L Ch R = 1 ,126016.6,874.9,874.9,874.9
BEGIN DESCRIPTION:
Town Creek 252.0
END DESCRIPTION:
#Sta/Elev= 30
  1157.8   83.46  1987.8   74.66  2047.8   76.46  2077.8   74.96  2227.8   75.74
  3017.8   69.81  3037.8   67.52  3057.8   68.48  3227.8   68.15  3257.8   65.46
  3277.8   67.54  3777.8   69.24  3797.8   70.28  4067.8   68.62    4325   69.39
  4447.8   66.32  4497.8   62.45  4527.8   65.87  4647.8   61.98  4757.8   61.12
  4947.8   62.08  4975.5   60.09 4976.55   57.09 5023.45   57.09  5024.5   60.09
    5320   62.95    5390   70.66    5480   89.14    5590   96.36    5653   98.28
#Mann= 4 , 1 , 0
 1157.80     0.2       0    4325    0.15       0  4975.5    0.05       0
  5024.5    0.15       0
Bank Sta=4975.50,5024.50
Exp/Cntr=0.3,0.1

Type RM Length L Ch R = 1 ,125141.7,1247.9,1247.9,1247.9
BEGIN DESCRIPTION:
Town Creek 250.0
END DESCRIPTION:
#Sta/Elev= 30
  1323.6   82.42  1603.6   76.01  1743.6   74.97  1753.6   73.41  1763.6   74.63
  2473.6   72.43  2773.6    67.6  2993.6   69.02  3143.6   68.05  3243.6   69.49
  3473.6   68.15  3623.6   70.09  3643.6   68.55  3803.6   70.75    3910   70.67
  4183.6   67.13  4253.6   68.97  4433.3   68.42  4453.3   69.66  4643.3   66.19
  4743.3   60.65  4803.3   61.32  4975.5   59.49 4976.55   56.49 5023.38   56.49
 5024.43   59.49  5033.3   72.36  5103.3   91.22  5183.3   97.02  5258.4   97.34
#Mann= 4 , 1 , 0
 1323.60     0.2       0    3910    0.15       0  4975.5    0.05       0
 5024.43    0.15       0
Bank Sta=4975.50,5024.43
Exp/Cntr=0.3,0.1

Type RM Length L Ch R = 1 ,123893.8,686.1,686.1,686.1
BEGIN DESCRIPTION:
Town Creek 248.0
END DESCRIPTION:
#Sta/Elev= 30
  1960.1   74.82  2600.1    70.6  2910.1   67.65  2930.1   66.06  2950.1   67.21
  3400.1   68.34  3420.1   66.71  3430.1   67.95  3650.1   67.07  3710.1   63.13
  3740.1   62.68  3840.1   65.41  3930.1   61.75  4180.1   62.53  4270.1   61.21
  4530.5   65.04  4570.5   63.29  4610.5   62.92  4630.5   61.01  4890.5   63.12
  4920.5   64.37  4960.5    63.9  4975.5   58.72 4976.55   55.72 5023.38   55.72
 5024.43   58.72  5080.5   66.42  5130.5   74.75  5230.5   85.62    5414   91.78
#Mann= 3 , 1 , 0
 1960.10    0.15       0  4975.5    0.05       0 5024.43    0.15       0
Bank Sta=4975.50,5024.43
Exp/Cntr=0.3,0.1

Type RM Length L Ch R = 1 ,123207.7,675.2,675.2,675.2
BEGIN DESCRIPTION:
Town Creek 246.0
END DESCRIPTION:
#Sta/Elev= 30
  2889.2   81.28  2899.2   80.29  2919.2   65.09  2929.2   64.32  2999.2   65.02
  3079.2   63.62  3559.2   64.46  3699.2   67.31  3759.2   66.12  3969.2   65.46
  4059.2   62.43  4159.2   64.08  4309.2    60.2  4359.2   62.41  4559.2   60.89
  4709.2   61.54  4729.2   60.51  4819.2   60.95  4929.2   62.84  4975.5   58.64
 4976.55   55.64 5023.45   55.64  5024.5   58.64  5214.3   61.93  5314.3   61.53
  5334.3   63.73  5434.3   69.48  5504.3   77.62  5584.3   91.49  5609.9   93.33
#Mann= 3 , 1 , 0
 2889.20    0.15       0  4975.5    0.05       0  5024.5    0.15       0
Bank Sta=4975.50,5024.50
Exp/Cntr=0.3,0.1

Type RM Length L Ch R = 1 ,122532.5,640.6,640.6,640.6
BEGIN DESCRIPTION:
Town Creek 245.0
END DESCRIPTION:
#Sta/Elev= 30
  3013.5    75.6  3373.5   64.32  3623.5   65.65  3673.5   63.07  3713.5   62.79
  3913.5   65.13  3983.5    62.6  4162.4    66.6  4212.4   65.65  4262.4   62.95
  4412.4   61.73  4452.4   60.01  4782.4   60.51  4812.4    59.4  4952.4   61.69
 4975.57   58.56 4976.62   55.56 5023.45   55.56  5024.5   58.56  5042.4    61.5
  5072.4   61.15  5121.2   62.76  5171.2   60.97  5271.2   60.24  5331.2   62.39
  5381.2   66.66  5451.2   75.69  5551.2   86.28  5601.2   89.86    5677   88.76
#Mann= 3 , 1 , 0
 3013.50    0.15       0 4975.57    0.05       0  5024.5    0.15       0
Bank Sta=4975.57,5024.50
Exp/Cntr=0.5,0.3
