--- White_Oak_Swamp_US_021220.prj (project) ---

Proj Title=White Oak Swamp US - Wilson County
Current Plan=p01
Default Exp/Contr=0.3,0.1
English Units
Geom File=g01
Flow File=f02
Flow File=f01
Plan File=p02
Plan File=p01
Y Axis Title=Elevation
X Axis Title(PF)=Main Channel Distance
X Axis Title(XS)=Station
BEGIN DESCRIPTION:
NEUSE RIVER BASIN
Little Contentnea Creek Sub-basin
WHITE OAK SWAMP
(Flood Hazard, Floodway) Model
Prepared by: Andrew J. Bonner   Date: 11/26/2002
Watershed Concepts
3333 Regency Pkwy
Cary, North Carolina 27511
END DESCRIPTION:
DSS Export Rating Curves= 0
DSS Export Rating Curve Sorted= 0
DSS Export Volume Flow Curves= 0
DXF OffsetX= 0
DXF OffsetY= 0
DXF ScaleX= 1
DXF ScaleY= 10

--- White_Oak_Swamp_US_021220.p01 (plan) ---

Plan Title=100 Year Single
Program Version=4.00
Short Identifier=100 Year Sin
Geom File=g01
Flow File=f01
Subcritical Flow
K Sum by GR= 0
Std Step Tol= 0.01
Critical Tol= 0.01
Num of Std Step Trials= 20
Max Error Tol= 0.3
Flow Tol Ratio= 0.001
Split Flow NTrial= 30
Split Flow Tol= 0.02
Split Flow Ratio= 0.02
Log Output Level= 0
Friction Slope Method= 1
Unsteady Friction Slope Method= 2
Unsteady Bridges Friction Slope Method= 1
Parabolic Critical Depth
Global Vel Dist= 0 , 0 , 0
Global Log Level= 0
CheckData=True
Encroach Param=-1 ,10,10, 2
Encroach River=White Oak US
Encroach Reach=Reach - 1
Encroach Node=38864.2
       4      .7
Encroach Node=38168.0
       4      .7
Encroach Node=37399.9
       4      .7
Encroach Node=37000.0
       4      .7
Encroach Node=36651.8
       4      .7
Encroach Node=35866.8
       4      .7
Encroach Node=35175.9
       4      .7
Encroach Node=34636.0
       4      .7
Encroach Node=33947.8
       4      .7
Encroach Node=33108.8
       4      .7
Encroach Node=32473.9
       4      .7
Encroach Node=31703.4
       4      .7
Encroach Node=31050.2
       4      .7
Encroach Node=30457.2
       4      .7
Encroach Node=29574.8
       4      .7
Encroach Node=28824.7
       4      .7
Encroach Node=28267.5
       4      .7
Encroach Node=27500.0
       4      .7
Encroach Node=26839.1
       4      .7
Encroach Node=26000.0
       4      .7
Encroach Node=25186.8
       4      .7
Encroach Node=24644.4
       4      .7
Encroach Node=24000.0
       4      .7
Encroach Node=23062.7
       4      .7
Encroach Node=22519.0
       1    4800    5230
Encroach Node=22473.0
       1    4800    5230
Encroach Node=21946.4
       4      .7
Encroach Node=21147.0
       4      .7
Encroach Node=20620.0
       4      .7
Encroach Node=19597.5
       4      .7
Encroach Node=18689.8
       4      .7
Encroach Node=17727.1
       4      .7
Encroach Node=16772.2
       4      .7
Encroach Node=15459.6
       4      .7
Encroach Node=14863.3
       4      .7
Encroach Node=13990.9
       4      .7
Encroach Node=13307.4
       4      .7
Encroach Node=12380.5
       1 4705.38 5255.38
Computation Interval=1HOUR
Output Interval=1HOUR
Run HTab= 0
Run UNet= 0
Run PostProcess= 0
Run WQNet= 0
UNET Theta= 1
UNET Theta Warmup= 1
UNET ZTol= 0.02
UNET ZSATol= 0.1
UNET MxIter= 20
UNET MaxInSteps= 20
UNET DtIC= 0
UNET DtMin= 0
UNET MaxCRTS= 20
UNET WFStab= 2
UNET SFStab= 1
UNET WFX= 1
UNET SFX= 1
UNET DSS MLevel= 4
UNET DZMax Abort= 100
UNET Convert EG Bridges=-1
UNET Use Existing IB Tables=-1
UNET Froude Reduction=False
UNET Froude Limit= 1
UNET Froude Power= 10
UNET Time Slicing=0,0, 5
Instantaneous Interval=1HOUR
DSS File=dss
Write IC File= 0
Echo Input=False
Echo Output=False
Write Detailed= 0
Detailed Automatic Start=False, 10
WQ ULTIMATE=-1
WQ Max Comp Step=1HOUR
WQ Output Interval=15MIN
WQ Output Selected Increments= 0
WQ Output face flow=0
WQ Output face velocity=0
WQ Output face area=0
WQ Output face dispersion=0
WQ Output cell volume=0
WQ Output cell surface area=0
WQ Output cell continuity=0
WQ Output face conc=0
WQ Output face dconc_dx=0
WQ Output face courant=0
WQ Output face peclet=0
WQ Output face adv mass=0
WQ Output face disp mass=0
WQ Output cell mass=0
WQ Output cell source sink temp=0
WQ Output cell source sink nsm=0
WQ Output MaxMinRange=-1
WQ Daily Max Min Mean=-1
WQ Daily Range=0
WQ Daily Time=0
WQ Create Restart=0
WQ Fixed Restart=0
WQ System Summary=False
Sorting and Armoring Iterations= 10
XS Update Threshold= 0.02
Hydraulics Update Threshold= 0.02
Energy Slope Method= 1
Volume Change Method= 0
XS Weighting Method= 0
Number of US Weighted Cross Sections= 1
Number of DS Weighted Cross Sections= 1
Upstream XS Weight=0.25
Main XS Weight=0.5
Downstream XS Weight=0.25
Number of DS XS's Weighted with US Boundary= 1
Upstream Boundary Weight= 1
Weight of XSs Associated with US Boundary= 0
Number of US XS's Weighted with DS Boundary= 1
Downstream Boundary Weight= 0.5
Weight of XSs Associated with DS Boundary= 0.5
Sediment Output Level= 4
Mass or Volume Output= 0
Output Increment Type= 1
Profile and TS Output Increment= 10
XS Output Flag= 0
XS Output Increment= 10
Disregard all LS=0
Disregard all Conn=0
Disregard all Breaches=0
Disregard all Pumps=0

--- White_Oak_Swamp_US_021220.p02 (plan) ---

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Plan Title=Multi_Profile
Short Identifier=Multi_Profile
Geom File=g01
Flow File=f02
Encroach Param=-1 ,0,0, 0
UNET ZSATol= 0.05
UNET MaxInSteps= 0
UNET Convert EG Bridges= 0

--- White_Oak_Swamp_US_021220.f01 (steady flow) ---

Flow Title= 100 Year Single
Program Version=4.00
Number of Profiles= 2
Profile Names=100-Year,AFW
River Rch & RM=White Oak US,Reach - 1       ,38864.2
    2262    2262
River Rch & RM=White Oak US,Reach - 1       ,35866.8
    3073    3073
River Rch & RM=White Oak US,Reach - 1       ,28824.7
    4105    4105
River Rch & RM=White Oak US,Reach - 1       ,24000
    4574    4574
River Rch & RM=White Oak US,Reach - 1       ,18689.8
    4863    4863
River Rch & RM=White Oak US,Reach - 1       ,15459.6
    5550    5550
River Rch & RM=White Oak US,Reach - 1       ,12380.5
    5550    5550
Boundary for River Rch & Prof#=White Oak US,Reach - 1       , 1
Up Type= 0
Dn Type= 1
Dn Known WS=82.4
Boundary for River Rch & Prof#=White Oak US,Reach - 1       , 2
Up Type= 0
Dn Type= 1
Dn Known WS=83.12
DSS Import GetInterval= 0
DSS Import GetPeak= 0
DSS Import FillOption= 0

--- White_Oak_Swamp_US_021220.f02 (steady flow) ---

Flow Title=Multi_Profile
Program Version=4.00
Number of Profiles= 7
Profile Names=10yr,25yr,50yr,500yr,100yr-10%,100yr-20%,100yr-35%
River Rch & RM=White Oak US,Reach - 1       ,38864.2
    1083    1497    1860    3399    2446    3135    3831
River Rch & RM=White Oak US,Reach - 1       ,35866.8
    1498    2055    2540    4573    3272    4194    5124
River Rch & RM=White Oak US,Reach - 1       ,28824.7
    2036    2770    3409    6053    4307    5519    6744
River Rch & RM=White Oak US,Reach - 1       ,24000.0
    2283    3097    3805    6720    4772    6115    7472
River Rch & RM=White Oak US,Reach - 1       ,18689.8
    2436    3299    4049    7131    5057    6481    7919
River Rch & RM=White Oak US,Reach - 1       ,15459.6
    2802    3781    4631    8103    5732    7347    8977
Boundary for River Rch & Prof#=White Oak US,Reach - 1       , 1
Up Type= 0
Dn Type= 1
Dn Known WS=79.65
Boundary for River Rch & Prof#=White Oak US,Reach - 1       , 2
Up Type= 0
Dn Type= 1
Dn Known WS=80.75
Boundary for River Rch & Prof#=White Oak US,Reach - 1       , 3
Up Type= 0
Dn Type= 1
Dn Known WS=81.57
Boundary for River Rch & Prof#=White Oak US,Reach - 1       , 4
Up Type= 0
Dn Type= 1
Dn Known WS=83.51
Boundary for River Rch & Prof#=White Oak US,Reach - 1       , 5
Up Type= 0
Dn Type= 1
Dn Known WS=82.54
Boundary for River Rch & Prof#=White Oak US,Reach - 1       , 6
Up Type= 0
Dn Type= 1
Dn Known WS=83.43
Boundary for River Rch & Prof#=White Oak US,Reach - 1       , 7
Up Type= 0
Dn Type= 1
Dn Known WS=83.34
DSS Import GetInterval= 0
DSS Import GetPeak= 0
DSS Import FillOption= 0

--- White_Oak_Swamp_US_021220.g01 (geometry) ---

Geom Title=Geom 01 by CodeH2 for Windows
Program Version=4.00

River Reach=White Oak US    ,Reach - 1
Reach XY= 30
       0.9268516       0.6648419       0.9012524       0.6540357
       0.8900229       0.6329288       0.8832645       0.6420784
       0.8276949       0.6118495       0.7986913       0.4932364
       0.8100077       0.4763874       0.8065709       0.4367375
       0.7656641       0.4027882       0.7387562       0.3351414
       0.6463855        0.319429       0.5818137        0.285768
       0.5510338       0.2333767        0.503358       0.2096701
       0.4639336       0.1629111        0.427129       0.1701148
       0.4239859       0.1504681       0.3901934       0.1282017
       0.3669543       0.1439458       0.3120185       0.1264983
       0.2863764       0.1337836       0.2706076       0.1634351
       0.2810947       0.1860697       0.2707586       0.2200966
       0.2477468       0.2299047       0.2286581        0.264536
        0.145094       0.2409698       0.0873217         0.26425
       0.0643269       0.2945611       0.0522485       0.2936169

Type RM Length L Ch R = 1 ,38864.2 ,696.2,696.2,696.2
BEGIN DESCRIPTION:
White Oak Swamp US 42.0
END DESCRIPTION:
XS GIS Cut Line= 3
            0.95       0.6503613       0.9268956       0.6648294
       0.8943499       0.6937496
#Sta/Elev= 27
  4535.1  102.58  4675.1   99.16  4695.1   96.78  4745.1    93.2  4765.1   92.49
  4805.1   93.08  4945.1   91.85  4965.1   90.89  4992.5   90.59  4994.5   86.59
  5005.6   86.59  5007.6   90.59  5009.2   91.52  5049.2   90.58  5119.2   91.44
  5139.2    90.9  5159.2   92.08  5169.2      92  5189.2   93.19  5219.2   93.62
  5239.2   93.18  5249.2    92.4  5259.2   92.63  5299.2   95.01  5329.2    95.4
  5659.2   99.81  5740.4   99.14
#Mann= 3 , 1 , 0
  4535.1     .14       0  4992.5    .047       0  5007.6     .14       0
Bank Sta=4992.5,5007.6
XS Rating Curve= 0 ,0
Exp/Cntr=0.3,0.1

Type RM Length L Ch R = 1 ,38168.0 ,768.1,768.1,768.1
BEGIN DESCRIPTION:
White Oak Swamp US 41.0
END DESCRIPTION:
XS GIS Cut Line= 3
       0.9207601       0.6258375       0.9028389       0.6475317
       0.8745422       0.6711122
#Sta/Elev= 25
  4522.1  100.81  4802.1   94.86  4842.1   92.07  4952.1   90.44  4982.1   91.11
  4992.1   90.72  4992.5   89.39  4994.5   85.39  5005.6   85.39  5007.6   89.39
  5011.2   90.15  5191.2   91.04  5201.2   90.79  5221.2   91.33  5251.2   91.01
  5281.2    91.8  5311.2   91.89  5361.2   93.05  5381.2   94.04  5421.2   97.85
  5441.2   98.63  5541.2   98.36  5561.2   99.03  5581.2    98.8  5628.3   99.47
#Mann= 3 , 1 , 0
  4522.1     .14       0  4992.5    .047       0  5007.6     .14       0
Bank Sta=4992.5,5007.6
XS Rating Curve= 0 ,0
Exp/Cntr=0.3,0.1

Type RM Length L Ch R = 1 ,37399.9 ,399.9,399.9,399.9
BEGIN DESCRIPTION:
White Oak Swamp US 40.0
END DESCRIPTION:
XS GIS Cut Line= 3
       0.8886905       0.6126324       0.8815215        0.639661
       0.8698261       0.6692258
#Sta/Elev= 30
    4409  103.34    4479  100.92    4529   93.63    4559   91.24  4601.1   90.01
  4611.1   89.12  4631.1   90.08  4681.1   90.33  4691.1   89.93  4771.1   90.72
  4821.1   89.95  4841.1   90.54  4981.1   89.86  4991.1   89.49  4992.5   88.95
  4994.5   84.95  5005.6   84.95  5007.6   88.95  5012.1   90.06  5032.1   89.84
  5122.1   91.14  5172.1   91.42  5182.1   91.02  5212.1   91.75  5232.1   93.02
  5252.1    93.7  5272.1    93.6  5282.1   94.56  5402.1   99.09  5543.4  100.11
#Mann= 3 , 1 , 0
    4409     .14       0  4992.5    .047       0  5007.6     .14       0
Bank Sta=4992.5,5007.6
XS Rating Curve= 0 ,0
Exp/Cntr=0.3,0.1

Type RM Length L Ch R = 1 ,37000.0 ,348.2,348.2,348.2
BEGIN DESCRIPTION:
White Oak Swamp US 39.0
END DESCRIPTION:
XS GIS Cut Line= 3
        0.873599       0.6060298       0.8675043       0.6256264
       0.8566209         0.66168
#Sta/Elev= 30
  4650.6   98.21  4690.6   96.11  4700.6   96.06  4740.6    93.7  4760.6   91.27
  4800.6   89.87  4840.6   90.04  4890.6   88.67  4920.6   89.46  4960.6   89.18
  4970.6   89.41  4992.4   88.55  4994.4   84.55  5005.6   84.55  5007.6   88.55
    5010   89.09    5160   89.89    5190   91.51    5200   92.33    5290   93.96
    5330   93.61    5340   94.41    5350   93.56    5380   94.81    5400   94.59
    5410   94.95    5500   96.07    5520   96.64    5630    98.4  5641.1   98.26
#Mann= 3 , 1 , 0
  4650.6     .14       0  4992.4    .047       0  5007.6     .14       0
Bank Sta=4992.4,5007.6
XS Rating Curve= 0 ,0
Exp/Cntr=0.3,0.1

Type RM Length L Ch R = 1 ,36651.8 ,785,785,785
BEGIN DESCRIPTION:
White Oak Swamp US 38.0
END DESCRIPTION:
XS GIS Cut Line= 3
       0.8603938       0.5947112       0.8506814       0.6237091
       0.8471887       0.6522478
#Sta/Elev= 28
  4476.6  101.72  4496.6  101.39  4536.6   98.79  4566.6   97.82  4586.6   96.14
  4646.6   93.88  4706.6   93.34  4736.6    91.6  4756.6   90.03  4796.6   89.88
  4816.6   89.22  4826.6   89.68  4866.6   89.24  4886.6   88.39  4986.6    89.5
  4992.4   88.29  4994.4   84.29  5005.5   84.29  5007.5   88.29  5027.2   89.22
  5077.2   88.61  5197.2   90.29  5207.2   90.19  5267.2   93.76  5317.2   94.59
  5377.2   96.79  5447.2   97.65  5486.7   96.98
#Mann= 3 , 1 , 0
  4476.6     .14       0  4992.4    .047       0  5007.5     .14       0
Bank Sta=4992.4,5007.5
XS Rating Curve= 0 ,0
Exp/Cntr=0.3,0.1

Type RM Length L Ch R = 1 ,35866.8 ,690.9,690.9,690.9
BEGIN DESCRIPTION:
White Oak Swamp US 37.0
END DESCRIPTION:
XS GIS Cut Line= 3
       0.8613371       0.5890518       0.8290578       0.5985407
       0.7953115       0.6060298
#Sta/Elev= 24
  4422.4  102.66  4472.4  100.83  4502.4  100.18  4542.4   97.67  4562.4   96.94
  4582.4   95.52  4742.4   92.34  4912.4   90.02  4932.4   89.05  4982.4   88.61
  4990.1   87.33  4992.1   83.33  5007.8   83.33  5009.8   87.33  5045.2   88.07
  5115.2   88.97  5145.2   89.03  5225.2   90.47  5245.2   90.12  5255.2   90.48
  5295.2   93.89  5375.2   96.35  5535.2   99.53  5583.7  100.74
#Mann= 3 , 1 , 0
  4422.4     .14       0  4990.1    .047       0  5009.8     .14       0
Bank Sta=4990.1,5009.8
XS Rating Curve= 0 ,0
Exp/Cntr=0.3,0.1

Type RM Length L Ch R = 1 ,35175.9 ,539.9,539.9,539.9
BEGIN DESCRIPTION:
White Oak Swamp US 36.0
END DESCRIPTION:
XS GIS Cut Line= 3
       0.8594506       0.5616984       0.8245514       0.5683009
       0.7868225       0.5871654
#Sta/Elev= 30
  4398.1  101.09  4498.1   99.04  4548.1   97.02  4618.1   95.44  4638.1   96.22
  4658.1   95.07  4758.1   95.04  4778.1   95.64  4798.1   94.93  4808.1   95.45
  4848.1      95  4908.1      90  4928.1   88.88  4948.1   88.77  4990.1   86.45
  4992.1   82.45  5007.9   82.45  5009.9   86.45  5022.8   87.95  5222.8   88.64
  5242.8   89.34  5272.8   89.07  5392.8   91.85  5422.8   92.98  5472.8   92.48
  5512.8   93.13  5542.8   94.11  5572.8   97.05  5602.8   98.43  5720.9  102.14
#Mann= 3 , 1 , 0
  4398.1     .14       0  4990.1    .047       0  5009.9     .14       0
Bank Sta=4990.1,5009.9
XS Rating Curve= 0 ,0
Exp/Cntr=0.3,0.1

Type RM Length L Ch R = 1 ,34636.0 ,688.2,688.2,688.2
BEGIN DESCRIPTION:
White Oak Swamp US 35.0
END DESCRIPTION:
XS GIS Cut Line= 3
       0.8641667       0.5418907        0.813106       0.5464314
       0.7792767       0.5503797
#Sta/Elev= 30
  4125.1   104.5  4215.1  101.89  4435.1    97.3  4745.1   94.57  4795.1   91.67
  4805.1   91.99  4825.1   90.29  4845.1   90.48  4865.1   89.31  4885.1    90.3
  4925.1    87.7  4935.1   88.13  4955.1   87.48  4975.1   88.33  4985.1   87.92
  4990.1    86.2  4992.1    82.2  5007.8    82.2  5009.8    86.2  5027.8   88.41
  5087.8   88.98  5157.8   88.36  5227.8   88.71  5257.8   87.77  5337.8   88.72
  5417.8   93.01  5477.8   94.07  5527.8   95.86  5557.8   98.51  5577.7    99.2
#Mann= 3 , 1 , 0
  4125.1     .14       0  4990.1    .047       0  5009.8     .14       0
Bank Sta=4990.1,5009.8
XS Rating Curve= 0 ,0
Exp/Cntr=0.3,0.1

Type RM Length L Ch R = 1 ,33947.8 ,839,839,839
BEGIN DESCRIPTION:
White Oak Swamp US 34.0
END DESCRIPTION:
XS GIS Cut Line= 3
       0.8575642        0.513594       0.8060163       0.5116919
       0.7613554       0.5107643
#Sta/Elev= 30
  4114.1   98.81  4184.1   97.02  4194.1   96.01  4204.1   94.13  4214.1   94.34
  4234.1   96.13  4314.1   96.41  4514.1   93.35  4744.1   91.19  4794.1   88.57
  4914.1   87.38  4934.1   86.33  4954.1   87.58  4990.1   86.07  4992.1   82.07
  5007.8   82.07  5009.8   86.07  5042.3   88.26  5172.3   88.17  5192.3   88.75
  5252.3   88.01  5272.3   89.34  5322.3   89.89  5412.3   92.41  5452.3   92.09
  5492.3   93.17  5552.3   92.35  5612.3   96.04  5682.3   94.83  5752.8   98.18
#Mann= 3 , 1 , 0
  4114.1     .14       0  4990.1    .047       0  5009.8     .14       0
Bank Sta=4990.1,5009.8
XS Rating Curve= 0 ,0
Exp/Cntr=0.3,0.1

Type RM Length L Ch R = 1 ,33108.8 ,634.9,634.9,634.9
BEGIN DESCRIPTION:
White Oak Swamp US 33.0
END DESCRIPTION:
XS GIS Cut Line= 3
       0.8424726       0.4720922       0.8099156        0.474471
        0.767958        0.471149
#Sta/Elev= 26
  4445.8   98.93  4535.8   97.38  4595.8   95.93  4665.8   91.41  4675.8   90.51
  4725.8   90.79  4755.8    89.7  4775.8   90.11  4925.8   87.66  4945.8   87.66
  4965.8   87.16  4975.8   87.34  4990.1   85.91  4992.1   81.91  5007.8   81.91
  5009.8   85.91  5011.6   87.11  5051.6   87.07  5071.6   86.25  5081.6   86.76
  5151.6   87.77  5191.6   89.52  5261.6   89.22  5681.6   97.48  5711.6   97.34
  5718.1   97.55
#Mann= 3 , 1 , 0
  4445.8     .14       0  4990.1    .047       0  5009.8     .14       0
Bank Sta=4990.1,5009.8
XS Rating Curve= 0 ,0
Exp/Cntr=0.3,0.1

Type RM Length L Ch R = 1 ,32473.9 ,770.5,770.5,770.5
BEGIN DESCRIPTION:
White Oak Swamp US 32.0
END DESCRIPTION:
XS GIS Cut Line= 3
       0.8254946       0.4400226        0.801914       0.4437955
       0.7689012       0.4532278
#Sta/Elev= 24
  4593.6   99.08  4653.6   96.91  4693.6   95.72  4723.6   92.14  4743.6   90.51
  4763.6   90.13  4773.6   89.53  4793.6   89.72  4833.6    87.1  4853.6   87.74
  4883.6   87.21  4983.6    86.9  4990.2   85.79  4992.2   81.79  5007.9   81.79
  5009.9   85.79  5010.2   87.35  5030.2   87.07  5050.2   88.12  5060.2   88.23
  5080.2   87.64  5170.2    90.2  5200.2   89.56  5584.7   98.35
#Mann= 3 , 1 , 0
  4593.6     .14       0  4990.2    .047       0  5009.9     .14       0
Bank Sta=4990.2,5009.9
XS Rating Curve= 0 ,0
Exp/Cntr=0.3,0.1

Type RM Length L Ch R = 1 ,31703.4 ,653.2,653.2,653.2
BEGIN DESCRIPTION:
White Oak Swamp US 31.0
END DESCRIPTION:
XS GIS Cut Line= 3
       0.7943682       0.4098395       0.7851017       0.4205893
       0.7622987       0.4466252
#Sta/Elev= 25
  4757.5   96.55  4817.5   92.39  4857.5      91  4877.5   89.37  4887.5   88.15
  4917.5   87.16  4987.5   87.37  4990.1   85.65  4992.1   81.65  5007.9   81.65
  5009.9   85.65  5029.1   87.28  5049.1   86.48  5069.1   86.68  5079.1   87.15
  5149.1   86.96  5219.1   89.45  5239.1   91.08  5249.1   91.51  5259.1   90.97
  5309.1   92.51  5359.1   92.53  5379.1      93  5399.1   92.82  5588.3   96.35
#Mann= 3 , 1 , 0
  4757.5     .14       0  4990.1    .047       0  5009.9     .14       0
Bank Sta=4990.1,5009.9
XS Rating Curve= 0 ,0
Exp/Cntr=0.3,0.1

Type RM Length L Ch R = 1 ,31050.2 ,593,593,593
BEGIN DESCRIPTION:
White Oak Swamp US 30.0
END DESCRIPTION:
XS GIS Cut Line= 3
       0.7839928       0.3919183       0.7666685        0.394003
       0.7198536       0.4145556
#Sta/Elev= 22
  4697.1   99.71  4737.1   97.92  4797.1   94.64  4857.1   92.79  4867.1   91.59
  4907.1   88.25  4947.1    86.6  4977.1   86.99  4987.1   86.85  4990.1   85.52
  4992.1   81.52  5007.9   81.52  5009.9   85.52  5144.2   87.11  5254.2   87.37
  5284.2   87.31  5294.2    88.1  5304.2   89.46  5324.2   90.75  5334.2   90.36
  5374.2   90.45  5864.6   98.96
#Mann= 3 , 1 , 0
  4697.1     .14       0  4990.1    .047       0  5009.9     .14       0
Bank Sta=4990.1,5009.9
XS Rating Curve= 0 ,0
Exp/Cntr=0.3,0.1

Type RM Length L Ch R = 1 ,30457.2 ,882.4,882.4,882.4
BEGIN DESCRIPTION:
White Oak Swamp US 29.0
END DESCRIPTION:
XS GIS Cut Line= 3
       0.7943682       0.3579622       0.7547529       0.3626784
       0.7028756       0.3928615
#Sta/Elev= 28
  4319.2  102.64  4539.2   97.78  4599.2   93.36  4619.2   92.76  4649.2   93.01
  4679.2   91.21  4729.2   90.74  4779.2   87.77  4799.2   86.18  4989.2   86.23
  4990.1   85.41  4992.1   81.41  5007.9   81.41  5009.9   85.41  5078.4   87.18
  5088.4   87.53  5138.4   86.44  5198.4   88.08  5248.4    88.6  5258.4    88.1
  5298.4   88.46  5388.4      90  5568.4   94.37  5838.4   94.47  5898.4      96
  5988.4    97.8  6008.4    97.8  6020.2   98.13
#Mann= 3 , 1 , 0
  4319.2     .14       0  4990.1    .047       0  5009.9     .14       0
Bank Sta=4990.1,5009.9
XS Rating Curve= 0 ,0
Exp/Cntr=0.3,0.1

Type RM Length L Ch R = 1 ,29574.8 ,750.1,750.1,750.1
BEGIN DESCRIPTION:
White Oak Swamp US 28.0
END DESCRIPTION:
XS GIS Cut Line= 3
       0.7368316       0.2919367       0.7236265       0.3306088
        0.700046        0.390975
#Sta/Elev= 30
  4315.9   96.63  4325.9   95.35  4355.9   96.57  4375.9   95.86  4415.9   96.73
  4455.9   93.29  4605.9   87.87  4675.9    86.4  4705.9   86.56  4725.9   85.75
  4775.9    86.2  4835.9   85.31  4845.9   85.91  4905.9   85.46  4975.9   86.07
  4985.9   85.76  4990.2   84.77  4992.2   80.77  5007.9   80.77  5009.9   84.77
  5011.6   85.42  5021.6   85.76  5081.6   84.92  5151.6   85.87  5161.6   85.43
  5291.6   88.54  5311.6   88.16  5371.6   89.23  5681.6   91.73    6115   98.05
#Mann= 3 , 1 , 0
  4315.9     .14       0  4990.2    .047       0  5009.9     .14       0
Bank Sta=4990.2,5009.9
XS Rating Curve= 0 ,0
Exp/Cntr=0.3,0.1

Type RM Length L Ch R = 1 ,28824.7 ,557.2,557.2,557.2
BEGIN DESCRIPTION:
White Oak Swamp US 27.0
END DESCRIPTION:
XS GIS Cut Line= 3
       0.6868408       0.2957095       0.6869094       0.3305502
       0.6755222       0.3805996
#Sta/Elev= 30
  4404.2   97.29  4454.2   87.26  4464.2   86.33  4494.2   85.48  4564.2   84.43
  4694.2   85.49  4704.2   84.81  4794.2   84.43  4854.2   85.33  4884.2   84.74
  4924.2      86  4986.7   84.72  4988.7   80.72  5011.4   80.72  5013.4   84.72
  5027.4   86.69  5087.4   85.49  5167.4   85.36  5217.4    86.1  5237.4   85.66
  5257.4   87.32  5337.4   89.11  5367.4   88.26  5557.4   93.49  5587.4   93.47
  5627.4   95.41  5667.4   94.99  5697.4   97.12  5837.4   100.7  5871.2  100.69
#Mann= 3 , 1 , 0
  4404.2     .14       0  4986.7    .047       0  5013.4     .14       0
Bank Sta=4986.7,5013.4
XS Rating Curve= 0 ,0
Exp/Cntr=0.3,0.1

Type RM Length L Ch R = 1 ,28267.5 ,767.5,767.5,767.5
BEGIN DESCRIPTION:
White Oak Swamp US 26.0
END DESCRIPTION:
XS GIS Cut Line= 3
       0.6651467       0.3008973       0.6589051       0.3181432
       0.6462823       0.3725822
#Sta/Elev= 30
  4686.5      95  4716.5   88.26  4756.5   86.15  4906.5   84.91  4976.5   85.18
  4986.6    84.1  4988.6    80.1  5011.4    80.1  5013.4    84.1  5268.7   85.41
  5308.7   84.71  5378.7   85.03  5478.7   84.46  5488.7   84.79  5518.7   86.74
  5538.7   87.42  5558.7   88.61  5618.7   89.56  5638.7   90.41  5658.7   90.37
  5698.7   91.69  5718.7   91.55  5738.7   92.12  5748.7   92.89  5758.7   94.15
  5788.7   95.42  5838.7   96.39  5848.7   96.23  5948.7   98.86  5950.1   98.94
#Mann= 3 , 1 , 0
  4686.5     .14       0  4986.6    .047       0  5013.4     .14       0
Bank Sta=4986.6,5013.4
XS Rating Curve= 0 ,0
Exp/Cntr=0.3,0.1

Type RM Length L Ch R = 1 ,27500.0 ,660.9,660.9,660.9
BEGIN DESCRIPTION:
White Oak Swamp US 25.0
END DESCRIPTION:
XS GIS Cut Line= 3
       0.6293042       0.2801464         0.62373       0.3093014
       0.6076101       0.3754119
#Sta/Elev= 30
  4494.7   99.35  4504.7   98.21  4524.7   96.71  4544.7   93.39  4584.7   91.19
  4594.7   91.11  4624.7   88.73  4634.7   87.42  4654.7   86.76  4674.7   85.24
  4734.7    83.9  4754.7   84.46  4774.7   83.69  4964.7   84.69  4986.7   83.89
  4988.7   79.89  5011.4   79.89  5013.4   83.89    5060   85.45    5200   85.65
    5210   85.18    5340   88.23    5370    88.5    5390   87.94    5460   89.28
    5500    91.9    5540   91.03    5910   94.43    6130   98.58  6158.5   99.54
#Mann= 3 , 1 , 0
  4494.7     .14       0  4986.7    .047       0  5013.4     .14       0
Bank Sta=4986.7,5013.4
XS Rating Curve= 0 ,0
Exp/Cntr=0.3,0.1

Type RM Length L Ch R = 1 ,26839.1 ,839.1,839.1,839.1
BEGIN DESCRIPTION:
White Oak Swamp US 24.0
END DESCRIPTION:
XS GIS Cut Line= 3
        0.611383        0.274487       0.5915529       0.2901389
       0.5538464       0.3263643
#Sta/Elev= 30
  4565.1  101.15  4585.1   96.77  4615.1   93.58  4705.1   89.25  4775.1   88.28
  4825.1   85.08  4845.1    84.5  4865.1   85.13  4945.1   84.79  4986.7   83.71
  4988.7   79.71  5011.4   79.71  5013.4   83.71  5135.2   84.95  5165.2   84.13
  5195.2   85.75  5265.2   85.12  5315.2   86.83  5395.2    86.6  5405.2   85.99
  5415.2   87.12  5435.2    87.2  5455.2   88.55  5665.2   90.78  5685.2   92.08
  5735.2   92.27  5745.2   92.63  5775.2    96.4  5815.2   95.39  5885.4   97.92
#Mann= 3 , 1 , 0
  4565.1     .14       0  4986.7    .047       0  5013.4     .14       0
Bank Sta=4986.7,5013.4
XS Rating Curve= 0 ,0
Exp/Cntr=0.3,0.1

Type RM Length L Ch R = 1 ,26000.0 ,813.2,813.2,813.2
BEGIN DESCRIPTION:
White Oak Swamp US 23.0
END DESCRIPTION:
XS GIS Cut Line= 3
       0.5868592       0.2282691       0.5638185       0.2538171
       0.5151743       0.2971244
#Sta/Elev= 30
  4414.3    99.1  4434.3   99.12  4444.3   98.78  4464.3   96.94  4514.3   91.04
  4534.3   89.86  4554.3   89.23  4564.3   88.53  4584.3   89.36  4594.3   87.11
  4604.3   85.35  4664.3   83.47  4674.3   83.74  4694.3   83.45  4704.3   83.72
  4874.3   83.72  4974.3   84.54  4986.6   83.48  4988.6   79.48  5011.4   79.48
  5013.4   83.48    5140   83.42    5290   85.08    5450   87.62    5570    87.8
    5600   87.09    5640   87.42    5680   90.99    6100   98.57  6108.8   99.01
#Mann= 3 , 1 , 0
  4414.3     .14       0  4986.6    .047       0  5013.4     .14       0
Bank Sta=4986.6,5013.4
XS Rating Curve= 0 ,0
Exp/Cntr=0.3,0.1

Type RM Length L Ch R = 1 ,25186.8 ,542.4,542.4,542.4
BEGIN DESCRIPTION:
White Oak Swamp US 22.0
END DESCRIPTION:
XS GIS Cut Line= 3
       0.5469228       0.2058142        0.530936       0.2249137
       0.4831047       0.2839193
#Sta/Elev= 30
  4571.8  101.04  4581.8  100.26  4591.8   97.86  4621.8   86.34  4641.8   85.68
  4671.8    83.4  4981.8   83.83  4986.6   82.68  4988.6   78.68  5011.4   78.68
  5013.4   82.68  5015.8   83.73  5105.8   84.41  5165.8   83.57  5185.8   83.93
  5315.8   83.78  5405.8   85.58  5425.8   85.42  5455.8   86.17  5515.8   86.03
  5675.8   88.46  5695.8    90.2  5705.8   90.69  5735.8   88.89  5775.8   89.21
  5795.8   90.19  5815.8   90.13  5835.8   89.85  6255.8   97.46    6289   98.45
#Mann= 3 , 1 , 0
  4571.8     .13       0  4986.6    .047       0  5013.4     .13       0
Bank Sta=4986.6,5013.4
XS Rating Curve= 0 ,0
Exp/Cntr=0.3,0.1

Type RM Length L Ch R = 1 ,24644.4 ,644.4,644.4,644.4
BEGIN DESCRIPTION:
White Oak Swamp US 21.0
END DESCRIPTION:
XS GIS Cut Line= 4
       0.5198904       0.1707325       0.5065988       0.2108547
       0.4939523       0.2388578       0.4793318       0.2697709
#Sta/Elev= 30
  4278.1   97.12  4348.1    84.1  4378.1   83.01  4448.1   83.42  4538.1      83
  4558.1   82.42  4578.1   82.87  4588.1   82.75  4598.1   83.21  4788.1   82.94
  4808.1   82.19  4938.1   83.17  4986.7   82.41  4988.7   78.41  5011.4   78.41
  5013.4   82.41  5027.7   83.87  5097.7   83.71  5257.7   85.48  5277.7   85.03
  5307.7   85.99  5337.7    85.7  5367.7   86.71  5457.7   86.99  5497.7   88.31
  5520.8   88.19  5830.8   91.98  5900.8    92.8  5930.8   94.02    6103   98.27
#Mann= 3 , 1 , 0
  4278.1     .13       0  4986.7    .047       0  5013.4     .13       0
Bank Sta=4986.7,5013.4
XS Rating Curve= 0 ,0
Exp/Cntr=0.3,0.1

Type RM Length L Ch R = 1 ,24000.0 ,937.3,937.3,937.3
BEGIN DESCRIPTION:
White Oak Swamp US 20.0
END DESCRIPTION:
XS GIS Cut Line= 3
       0.4981963       0.1480952       0.4846896        0.185876
       0.4566945       0.2650548
#Sta/Elev= 30
  4316.9   98.39  4356.9   94.71  4426.9   84.21  4486.9   82.24  4516.9   83.11
  4606.9   82.31  4736.9   82.92  4756.9   82.11  4806.9   83.12  4936.9   82.51
  4966.9   83.12  4976.9   83.02  4984.8   81.61  4986.8   77.61  5013.1   77.61
  5015.1   81.61    5020   82.27    5210   82.99    5270   82.36    5400   82.43
    5520    85.4    5680   86.19    5700   85.44    5720   86.59    5750   86.04
    5980   90.65    6170   92.07    6220   93.44    6250   92.93  6429.8    98.1
#Mann= 3 , 1 , 0
  4316.9     .13       0  4984.8    .047       0  5015.1     .13       0
Bank Sta=4984.8,5015.1
XS Rating Curve= 0 ,0
Exp/Cntr=0.3,0.1

Type RM Length L Ch R = 1 ,23062.7 ,543.7,543.7,543.7
BEGIN DESCRIPTION:
White Oak Swamp US 19.0
END DESCRIPTION:
XS GIS Cut Line= 3
       0.4614106       0.1226282       0.4486955       0.1653602
        0.420852       0.2622251
#Sta/Elev= 30
  4241.8   97.36  4501.8   91.11  4631.8   88.54  4651.8   88.51  4691.8   87.09
  4711.8    85.8  4731.8   85.78  4791.8   84.21  4971.8   82.43  4984.8   81.44
  4986.8   77.44  5013.1   77.44  5015.1   81.44  5020.8   82.72  5110.8   81.76
  5150.8   82.77  5170.8   82.08  5260.8   82.87  5640.8   82.84  5650.8   82.36
  5670.8   82.68  5680.8   82.11  5830.8   83.66  5840.8   85.07  5880.8   86.58
  5910.8   86.41  5930.8   87.51  6100.8    88.5  6440.8    92.8  6716.7   97.28
#Mann= 3 , 1 , 0
  4241.8     .13       0  4984.8    .047       0  5015.1     .13       0
Bank Sta=4984.8,5015.1
XS Rating Curve= 0 ,0
Exp/Cntr=0.5,0.3

Type RM Length L Ch R = 1 ,22519.0 ,46,46,46
BEGIN DESCRIPTION:
Upstream Section of Bridge/Culvert/Weir
END DESCRIPTION:
XS GIS Cut Line= 5
       0.4404084       0.1258995        0.423672       0.1670279
       0.4184912       0.1768383       0.4156713       0.1910222
       0.4135713       0.2213275
#Sta/Elev= 30
  3981.5   98.36  4051.5   96.66  4081.5   94.35  4111.5    94.7  4241.5   91.36
  4261.5   89.92  4361.5   89.28  4421.5   86.25  4581.5    83.8  4601.5   82.69
  4671.5   82.46  4751.5   83.64  4821.5   82.96  4911.5   83.48  4941.5   81.94
  4971.5    82.4  4972.5   79.91    4985   77.11    5015   77.11  5027.5   79.91
    5041   82.26    5111   81.83    5391   83.57    5421   82.94  5539.7   85.31
  5629.7   84.34  5719.7   85.62  5779.7   88.11  5799.7   87.65  6316.6   92.41
#Mann= 3 , 1 , 0
  3981.5     .13       0  4972.5    .047       0  5027.5     .13       0
#XS Ineff= 2 , 0
       0    4947    84.5    5053       0    84.5
Permanent Ineff=
       F       F
Bank Sta=4972.5,5027.5
XS Rating Curve= 0 ,0
Exp/Cntr=0.5,0.3

Type RM Length L Ch R = 3 ,22496.0 ,,,
BEGIN DESCRIPTION:
Gardners School Rd-TOR
Structure ID: Gardners School Rd
Approximate Survey Structure
END DESCRIPTION:
Bridge Culvert--1,0,-1,-1, 0
Deck Dist Width WeirC Skew NumUp NumDn MinLoCord MaxHiCord MaxSubmerge Is_Ogee
10,26,2.6,0, 53, 53, , , 0.95, 0, 1,1,,
  3981.5  4051.5  4081.5  4111.5  4211.5  4241.5  4251.5  4261.5  4301.5  4321.5
  4331.5  4361.5  4371.5  4421.5  4470.3  4490.3  4521.5  4581.5  4601.5  4621.5
  4671.5  4751.5  4811.5  4821.5  4891.5  4911.5  4920.3  4941.5 4956.91    4957
 5042.89    5043    5091    5111    5341    5391    5421  5431.3  5509.7  5539.7
  5569.7  5609.7  5629.7  5659.7  5679.7  5699.7  5719.7  5779.7  5799.7  6089.7
  6189.7  6209.7  6316.6
   98.35   96.65   94.34   94.69   91.59   91.35   90.84   89.91   90.04   89.43
   89.92   89.27   88.25   86.24      86   85.54   85.52   85.48   85.45   85.42
   85.35   85.27   85.15   85.13   84.99   84.95   84.93   84.94   84.94   84.94
   84.99   84.99   85.02   85.04    85.1   85.11   85.33   85.42   85.57   85.63
   85.69   85.75   85.76   85.79   85.87   86.02    86.2    88.1   87.64   90.58
   91.05   91.65    92.4
   98.35   96.65   94.34   94.69   91.59   91.35   90.84   89.91   90.04   89.43
   89.92   89.27   88.25   86.24   85.41   85.07   84.54   83.79   82.68   83.15
   82.45   83.63   83.37   82.95   82.89   83.47   83.02   81.93   82.17   83.54
   83.59   82.25   82.29   81.82   83.13   83.56   82.93   83.13   84.62    85.3
    84.7   84.82   84.33   85.32   84.73   85.75   85.61    88.1   87.64   90.58
   91.05   91.65    92.4
  3981.5  4051.5  4081.5  4111.5  4211.5  4241.5  4251.5  4261.5  4301.5  4321.5
  4331.5  4361.5  4371.5  4421.5  4470.3  4490.3  4521.5  4581.5  4601.5  4621.5
  4671.5  4751.5  4811.5  4821.5  4891.5  4911.5  4920.3  4941.5 4956.91    4957
 5042.89    5043    5091    5111    5341    5391    5421  5431.3  5509.7  5539.7
  5569.7  5609.7  5629.7  5659.7  5679.7  5699.7  5719.7  5779.7  5799.7  6089.7
  6189.7  6209.7  6316.6
   98.25   96.55   94.24   94.59   91.49   91.26   90.75   89.82   89.95   89.34
   89.83   89.18   88.16   86.23      86   85.54   85.52   85.48   85.45   85.42
   85.35   85.27   85.15   85.13   84.99   84.95   84.93   84.94   84.94   84.94
   84.99   84.99   85.02   85.04    85.1   85.11   85.33   85.42   85.57   85.63
   85.69   85.75   85.76   85.79   85.87   86.02    86.2   88.01   87.55   90.48
   90.95   91.55    92.3
   98.15   96.45   94.14   94.49   91.39   91.15   90.64   89.71   89.84   89.23
   89.72   89.07   88.05   86.04   85.21   84.87   84.34   83.59   82.48   82.95
   82.25   83.43   83.17   82.75   82.69   83.27   82.82   81.73   81.97   83.34
   83.39   82.05   82.09   81.62   82.93   83.36   82.73   82.93   84.42    85.1
    84.5   84.62   84.13   85.12   84.53   85.55   85.41    87.9   87.44   90.38
   90.85   91.45    92.2
Pier Skew, UpSta & Num, DnSta & Num=  ,4974.5, 2 ,4974.5, 2 , 0 , 0 , 0 ,,
       1       1
   78.34   84.55
       1       1
   78.14   84.35
Pier Skew, UpSta & Num, DnSta & Num=  ,4991.5, 2 ,4991.5, 2 , 0 , 0 , 0 ,,
       1       1
    76.1   84.55
       1       1
    75.9   84.35
Pier Skew, UpSta & Num, DnSta & Num=  ,5008.5, 2 ,5008.5, 2 , 0 , 0 , 0 ,,
       1       1
    76.1   84.57
       1       1
    75.9   84.37
Pier Skew, UpSta & Num, DnSta & Num=  ,5025.5, 2 ,5025.5, 2 , 0 , 0 , 0 ,,
       1       1
   78.34   84.58
       1       1
   78.14   84.38
Abutment Skew #Up #Dn= , 2 , 2
  4956.8    4966
   83.54   82.31
  4956.8    4966
   83.34   82.11
Abutment Skew #Up #Dn= , 2 , 2
    5034 5043.09
   81.03   83.59
    5034 5043.09
   80.83   83.39
BR Coef= 1 , 1 , 0 ,1.25, 0 ,,,0.8,0,2,0,
WSPro=,,,, 1 ,,,, 0 ,,,, 0 ,,,,-1 ,-1 ,-1 , 0 , 0 , 0 , 0 , 0
BR U #Sta/Elev= 80
  3981.5   98.35  4051.5   96.65  4081.5   94.34  4111.5   94.69  4211.5   91.59
  4240.3   91.36  4241.5   91.35  4251.5   90.84  4261.5   89.91  4280.3   89.97
  4300.3   90.04  4301.5   90.04  4310.3   89.77  4321.5   89.43  4331.5   89.92
  4350.3   89.51  4361.5   89.27  4370.3   88.37  4371.5   88.25  4421.5   86.24
  4470.3   85.41  4490.3   85.07  4521.5   84.54  4540.3   84.31  4580.3   83.81
  4581.5   83.79  4601.5   82.68  4621.5   83.15  4671.5   82.45  4690.3   82.73
  4751.5   83.63  4760.3   83.59  4811.5   83.37  4821.5   82.95  4891.5   82.89
  4911.5   83.47  4920.3   83.02  4941.5   81.93 4956.91   82.17    4957   82.17
    4966   82.31  4971.5   82.39  4972.5    79.9  4980.3   78.15    4985    77.1
    5015    77.1  5027.5    79.9    5034   81.03    5041   82.25 5042.89   82.25
    5043   82.25    5091   82.29    5111   81.82  5195.1    82.3    5341   83.13
    5391   83.56  5395.1   83.47    5421   82.93  5431.3   83.13  5509.7   84.62
  5539.7    85.3  5569.7    84.7  5591.3   84.76  5609.7   84.82  5629.7   84.33
  5659.7   85.32  5671.3   84.98  5679.7   84.73  5699.7   85.75  5711.3   85.67
  5719.7   85.61  5779.7    88.1  5791.3   87.83  5799.7   87.64  5891.3   88.57
  5931.3   88.97  6089.7   90.58  6189.7   91.05  6209.7   91.65  6316.6    92.4
BR U #Mann= 3
  3981.5     .13  4972.5    .047  5027.5     .13
BR U Banks=4972.5,5027.5
BR D #Sta/Elev= 80
  3981.5   98.15  4051.5   96.45  4081.5   94.14  4111.5   94.49  4211.5   91.39
  4240.3   91.16  4241.5   91.15  4251.5   90.64  4261.5   89.71  4280.3   89.77
  4300.3   89.84  4301.5   89.84  4310.3   89.57  4321.5   89.23  4331.5   89.72
  4350.3   89.31  4361.5   89.07  4370.3   88.17  4371.5   88.05  4421.5   86.04
  4470.3   85.21  4490.3   84.87  4521.5   84.34  4540.3   84.11  4580.3   83.61
  4581.5   83.59  4601.5   82.48  4621.5   82.95  4671.5   82.25  4690.3   82.53
  4751.5   83.43  4760.3   83.39  4811.5   83.17  4821.5   82.75  4891.5   82.69
  4911.5   83.27  4920.3   82.82  4941.5   81.73 4956.91   81.97    4957   81.97
    4966   82.11  4971.5   82.19  4972.5    79.7  4980.3   77.95    4985    76.9
    5015    76.9  5027.5    79.7    5034   80.83    5041   82.05 5042.89   82.05
    5043   82.05    5091   82.09    5111   81.62  5195.1    82.1    5341   82.93
    5391   83.36  5395.1   83.27    5421   82.73  5431.3   82.93  5509.7   84.42
  5539.7    85.1  5569.7    84.5  5591.3   84.56  5609.7   84.62  5629.7   84.13
  5659.7   85.12  5671.3   84.78  5679.7   84.53  5699.7   85.55  5711.3   85.47
  5719.7   85.41  5779.7    87.9  5791.3   87.63  5799.7   87.44  5891.3   88.37
  5931.3   88.77  6089.7   90.38  6189.7   90.85  6209.7   91.45  6316.6    92.2
BR D #Mann= 3
  3981.5     .13  4972.5    .047  5027.5     .13
BR D Banks=4972.5,5027.5
BC Design=,, 0 ,, 0 ,,,,,,
BC HTab HWMax=98.36
BC Use User HTab Curves=0
BC User HTab FreeFlow(D)= 0

Type RM Length L Ch R = 1 ,22473.0 ,526.6,526.6,526.6
BEGIN DESCRIPTION:
Downstream Section of Bridge/Culvert/Weir
END DESCRIPTION:
XS GIS Cut Line= 5
       0.4379917       0.1246911       0.4212553       0.1658195
       0.4160745         0.17563       0.4132546       0.1898138
       0.4111547       0.2201192
#Sta/Elev= 30
  3981.5   98.15  4051.5   96.45  4081.5   94.14  4111.5   94.49  4241.5   91.15
  4261.5   89.71  4361.5   89.07  4421.5   86.04  4581.5   83.59  4601.5   82.48
  4671.5   82.25  4751.5   83.43  4821.5   82.75  4911.5   83.27  4941.5   81.73
  4971.5   82.19  4972.5    79.7    4985    76.9    5015    76.9  5027.5    79.7
    5041   82.05    5111   81.62    5391   83.36    5421   82.73  5539.7    85.1
  5629.7   84.13  5719.7   85.41  5779.7    87.9  5799.7   87.44  6316.6    92.2
#Mann= 3 , 1 , 0
  3981.5     .13       0  4972.5    .047       0  5027.5     .13       0
#XS Ineff= 2 , 0
       0    4947    84.5    5053       0    84.5
Permanent Ineff=
       F       F
Bank Sta=4972.5,5027.5
XS Rating Curve= 0 ,0
Exp/Cntr=0.5,0.3

Type RM Length L Ch R = 1 ,21946.4 ,799.4,799.4,799.4
BEGIN DESCRIPTION:
White Oak Swamp US 18.0
END DESCRIPTION:
XS GIS Cut Line= 3
       0.4236817       0.1169688        0.413956       0.1433822
       0.3708612        0.232042
#Sta/Elev= 30
  4523.9   99.82  4553.9   94.45  4573.9   94.19  4603.9   92.55  4663.9    88.5
  4693.9   88.61  4723.9   84.24  4733.9   82.38  4793.9   81.32  4984.9    80.7
  4986.9    76.7  5013.2    76.7  5015.2    80.7  5143.1   81.92  5183.1   83.62
  5273.1   82.25  5593.1   82.01  5663.1   82.66  5683.1   82.07  5703.1   82.36
  5823.1   85.95  5863.1   85.27  6013.1   88.03  6193.1   89.59  6443.1   91.39
  6453.1   91.76  6463.1   91.61  6493.1   92.33  6623.1   94.35  6681.4   95.98
#Mann= 3 , 1 , 0
  4523.9     .13       0  4984.9    .047       0  5015.2     .13       0
Bank Sta=4984.9,5015.2
XS Rating Curve= 0 ,0
Exp/Cntr=0.3,0.1

Type RM Length L Ch R = 1 ,21147.0 ,527,527,527
BEGIN DESCRIPTION:
White Oak Swamp US 17.0
END DESCRIPTION:
XS GIS Cut Line= 4
       0.3831231       0.0877289       0.3802934       0.1377197
       0.3755773       0.1858241       0.3680315       0.2216666
#Sta/Elev= 30
  4143.7   99.87  4193.7   98.33  4223.7   93.67  4243.7   92.73  4283.7   86.08
  4313.7   84.18  4433.7    84.6  4713.7   80.74  4743.7   81.71  4973.7   81.39
  4984.9   80.41  4986.9   76.41  5013.2   76.41  5015.2   80.41  5116.1   81.75
  5206.1   81.77  5256.1   80.41  5296.1   81.78  5446.1   81.08  5456.1    82.4
  5566.1   81.43  5606.1   82.93  5626.1   81.69  5656.1   81.75  5736.1   86.17
  5766.1    86.5    5839   91.18    5919   90.12    6099   90.49  6442.6   94.64
#Mann= 3 , 1 , 0
  4143.7     .13       0  4984.9    .047       0  5015.2     .13       0
Bank Sta=4984.9,5015.2
XS Rating Curve= 0 ,0
Exp/Cntr=0.3,0.1

Type RM Length L Ch R = 1 ,20620.0 ,1022.5,1022.5,1022.5
BEGIN DESCRIPTION:
White Oak Swamp US 16.0
END DESCRIPTION:
XS GIS Cut Line= 3
       0.3510535       0.0613187       0.3562448       0.1341612
       0.3585993       0.2178937
#Sta/Elev= 30
  3746.7   96.41  3896.7   91.53  3956.7   91.37  4176.7   86.36  4296.7   85.07
  4326.7   83.07  4346.7   83.73  4496.7   82.18  4526.7    80.5  4566.7   82.27
  4606.7   80.88  4736.7   82.11  4796.7   80.65  4866.7   81.68  4984.9   80.35
  4986.9   76.35  5013.2   76.35  5015.2   80.35    5020    81.4    5090   80.73
    5140   82.12    5270   80.48    5440   80.76    5460   81.77    5790   81.64
    5900   86.72    5910   86.25    5980   90.12    6320   93.82  6416.1   96.17
#Mann= 3 , 1 , 0
  3746.7     .13       0  4984.9    .047       0  5015.2     .13       0
Bank Sta=4984.9,5015.2
XS Rating Curve= 0 ,0
Exp/Cntr=0.3,0.1

Type RM Length L Ch R = 1 ,19597.5 ,907.7,907.7,907.7
BEGIN DESCRIPTION:
White Oak Swamp US 15.0
END DESCRIPTION:
XS GIS Cut Line= 3
       0.2859711            0.05       0.3097375       0.1270759
       0.3382967       0.2086457
#Sta/Elev= 30
  3630.9  104.18  3680.9   98.44  3710.9   92.42  3780.9   82.55  3970.9   81.91
  4174.9   82.46  4410.9   80.97  4430.9   80.19  4440.9    80.9  4720.9   80.63
  4810.9   81.46  4850.9   80.77  4950.9   81.35  4984.9   80.22  4986.9   76.22
  5013.2   76.22  5015.2   80.22  5044.1   81.34  5104.1   80.21  5134.1   80.97
  5224.1   80.58  5284.1   82.27  5344.1   80.85  5504.1   80.62  5554.1   82.87
  5734.1   83.97  5924.1   87.63  6324.1   88.14  6354.1   89.61  6475.4   89.84
#Mann= 4 , 1 , 0
  3630.9      10       0  4174.9     .14       0  4984.9    .047       0
  5015.2     .14       0
Bank Sta=4984.9,5015.2
XS Rating Curve= 0 ,0
Exp/Cntr=0.3,0.1

Type RM Length L Ch R = 1 ,18689.8 ,962.7,962.7,962.7
BEGIN DESCRIPTION:
White Oak Swamp US 14.0
END DESCRIPTION:
XS GIS Cut Line= 3
       0.2463558       0.1358333       0.2727863       0.1548015
       0.3265297       0.2122343
#Sta/Elev= 30
  4451.5   94.54  4541.5   92.85  4621.5   88.91  4641.5   88.52  4661.5   87.06
  4691.5   86.02  4701.5   86.33  4731.5   84.68  4983.7   79.17  4985.7   75.17
  5014.3   75.17  5016.3   79.17  5025.4   80.01  5055.4   79.43  5145.4   80.39
  5175.4   79.01  5265.4    79.1  5305.4    80.3  5315.4   79.72  5385.4   80.57
  5585.4   81.02  5685.4   79.17  5705.4   80.89  5745.4   81.44  5795.4   80.96
  5835.4   82.23  5865.4   85.87  5905.4   86.81  6055.4   88.96  6344.5   90.96
#Mann= 3 , 1 , 0
  4451.5     .14       0  4983.7    .047       0  5016.3     .14       0
Bank Sta=4983.7,5016.3
XS Rating Curve= 0 ,0
Exp/Cntr=0.3,0.1

Type RM Length L Ch R = 1 ,17727.1 ,954.9,954.9,954.9
BEGIN DESCRIPTION:
White Oak Swamp US 13.0
END DESCRIPTION:
XS GIS Cut Line= 3
       0.2265481       0.1537545       0.2696807       0.1962004
        0.298233       0.2292123
#Sta/Elev= 30
  3963.1   93.81  4003.1   93.26  4073.1    87.6  4103.1   87.17  4153.1   82.15
  4323.1   78.68  4373.1   79.93  4523.1   79.61  4563.1    78.3  4603.1   79.24
  4683.1   78.29  4783.1   79.75  4883.1   78.69  4933.1   79.62  4983.7   77.96
  4985.7   73.96  5014.3   73.96  5016.3   77.96  5043.4    79.1  5143.4   79.78
  5233.4   78.15  5293.4   79.77  5333.4   78.87  5493.4   80.32  5503.4   79.02
  5563.4   79.02  5593.4   80.86  5623.4   85.82  5693.4   92.82  5736.4   95.06
#Mann= 3 , 1 , 0
  3963.1     .14       0  4983.7    .047       0  5016.3     .14       0
Bank Sta=4983.7,5016.3
XS Rating Curve= 0 ,0
Exp/Cntr=0.3,0.1

Type RM Length L Ch R = 1 ,16772.2 ,1312.6,1312.6,1312.6
BEGIN DESCRIPTION:
White Oak Swamp US 12.0
END DESCRIPTION:
XS GIS Cut Line= 3
       0.2086269       0.1679029       0.2491206        0.228813
       0.2963466       0.2820328
#Sta/Elev= 30
  3757.5   93.07  3787.5   92.34  3847.5   87.29  3897.5   85.55  3917.5   85.83
  4017.5   83.34  4047.5   83.85  4087.5   82.21  4317.5   80.87  4487.5   82.25
  4597.5   80.63  4617.5   81.27  4697.5   78.72  4847.5   79.87  4917.5   78.15
  4983.7   77.89  4985.7   73.89  5014.3   73.89  5016.3   77.89  5032.7   78.73
  5212.7   77.93  5242.7   78.95  5592.7   78.31  5622.7   79.79  5672.7   84.19
  5692.7   83.93  5722.7   86.52  5872.7   86.27  6132.7   91.84  6214.1   92.09
#Mann= 3 , 1 , 0
  3757.5     .14       0  4983.7    .047       0  5016.3     .14       0
Bank Sta=4983.7,5016.3
XS Rating Curve= 0 ,0
Exp/Cntr=0.3,0.1

Type RM Length L Ch R = 1 ,15459.6 ,596.3,596.3,596.3
BEGIN DESCRIPTION:
White Oak Swamp US 11.0
END DESCRIPTION:
XS GIS Cut Line= 3
       0.1911225       0.1933899       0.1994927       0.2596532
        0.200994       0.3414615
#Sta/Elev= 30
  3863.8   91.42  3943.8   90.76  3953.8   89.81  3973.8   84.41  4003.8   80.59
  4033.8   78.59  4073.8    77.9  4173.8   77.02  4303.8   78.02  4373.8   76.63
  4613.8   77.97  4633.8   76.78  4743.8   76.75  4773.8   78.27  4843.8   78.65
  4913.8   77.22  4973.8   78.08  4980.8   76.11  4982.8   72.11  5017.2   72.11
  5019.2   76.11  5030.9   77.55  5100.9   77.96  5130.9   76.97  5310.9   78.17
  5630.9   77.17  5830.9    78.7  5950.9   81.87  6030.9   81.64  6393.9   89.05
#Mann= 3 , 1 , 0
  3863.8     .14       0  4980.8    .047       0  5019.2     .14       0
Bank Sta=4980.8,5019.2
XS Rating Curve= 0 ,0
Exp/Cntr=0.3,0.1

Type RM Length L Ch R = 1 ,14863.3 ,872.4,872.4,872.4
BEGIN DESCRIPTION:
White Oak Swamp US 10.0
END DESCRIPTION:
XS GIS Cut Line= 3
       0.1642954       0.1952563        0.167979       0.2495149
       0.1737276       0.3367397
#Sta/Elev= 30
  4075.1   91.17  4165.1   90.21  4295.1   84.42  4325.1   83.79  4395.1   79.08
  4475.1    76.5  4535.1   76.13  4555.1    77.3  4785.1   76.94  4975.1   76.43
  4980.8   75.34  4982.8   71.34  5017.2   71.34  5019.2   75.34    5031   77.47
    5161   77.92    5201    79.3    5251   78.93    5311   75.93    5431   78.83
    5511   78.77    5561   77.22    5601   78.08    5641   77.12  5749.9   78.78
    5811   77.84    5841    79.2    5871   79.35    5891    80.6  6489.2   89.74
#Mann= 4 , 1 , 0
  4075.1     .14       0  4980.8    .047       0  5019.2     .14       0
  5749.9      10       0
Bank Sta=4980.8,5019.2
XS Rating Curve= 0 ,0
Exp/Cntr=0.3,0.1

Type RM Length L Ch R = 1 ,13990.9 ,683.5,683.5,683.5
BEGIN DESCRIPTION:
White Oak Swamp US 9.0
END DESCRIPTION:
XS GIS Cut Line= 3
       0.1256233        0.198086       0.1231721       0.2489478
        0.116191       0.3527745
#Sta/Elev= 30
  4131.9   83.95  4161.9   79.53  4201.9    79.5  4251.9   77.38  4291.9   79.11
  4411.9   77.21  4811.9   77.28  4861.9   76.07  4971.9   76.29  4980.8    75.2
  4982.8    71.2  5017.2    71.2  5019.2    75.2  5048.8   76.52  5088.8   75.77
  5278.8   77.14  5308.8   76.01  5478.8   75.58  5538.8   77.68  5688.8   75.68
  5948.8   76.74  5978.8   75.79  6079.9   79.58  6228.8   78.94  6328.8   76.78
  6398.8   79.66  6618.8   77.65  6688.8   81.05  6738.8      86  6770.4   90.54
#Mann= 4 , 1 , 0
  4131.9     .14       0  4980.8    .047       0  5019.2     .14       0
  6079.9      10       0
Bank Sta=4980.8,5019.2
XS Rating Curve= 0 ,0
Exp/Cntr=0.3,0.1

Type RM Length L Ch R = 1 ,13307.4 ,926.9,926.9,926.9
BEGIN DESCRIPTION:
White Oak Swamp US 8.0
END DESCRIPTION:
XS GIS Cut Line= 3
       0.0878944       0.2273259       0.0897087       0.2639779
       0.0926105       0.3499449
#Sta/Elev= 30
  4370.6   88.38  4530.6   82.69  4810.6   78.71  4890.6   76.57  4950.6   76.53
  4980.8   74.77  4982.8   70.77  5017.2   70.77  5019.2   74.77  5035.4   76.55
  5145.4   75.67  5195.4   76.18  5235.4   75.12  5275.4   76.32  5345.4   75.28
  5465.4   76.34  5495.4   75.16  5505.4   75.93  5555.4   75.47  5585.4   76.92
  5615.4   75.99  5695.4      78  5769.9   78.58  5845.4   77.84  5875.4   78.47
  5925.4    76.5  5975.4   76.07  6075.4   81.33  6165.4   81.59  6459.8   88.54
#Mann= 4 , 1 , 0
  4370.6     .14       0  4980.8    .047       0  5019.2     .14       0
  5769.9      10       0
Bank Sta=4980.8,5019.2
XS Rating Curve= 0 ,0
Exp/Cntr=0.3,0.1

Type RM Length L Ch R = 1 ,12380.5 ,0,0,0
BEGIN DESCRIPTION:
White Oak Swamp US 7.8 (Tie-in to new DTL STUDY)
END DESCRIPTION:
XS GIS Cut Line= 6
       0.0643138       0.2141208       0.0522458       0.2936181
       0.0503208        0.305168            0.05       0.3340426
       0.0564166       0.3452716       0.0634748       0.3494424
#Sta/Elev= 30
 3655.38   88.25 3715.25   84.91 3814.91   77.38 3881.38   77.27 3894.83   76.21
 3912.46   77.38 4036.89   75.65 4101.27   76.84 4165.38   75.53 4298.41   75.22
 4533.38   76.32 4599.01   76.14 4616.73   74.96 4717.66   76.55  4985.3   75.18
    4989   74.98 4992.83   70.56 5007.07   70.59  5010.4   74.62 5021.55   75.51
 5170.63   75.56 5287.05   79.55 5353.94   79.55 5427.12    76.8  5499.8    77.7
 5526.82   79.21 5597.02   79.03 5727.81   81.69 5983.08   82.54 6020.19   84.44
#Mann= 7 ,-1 , 0
 3655.38    .045       0 3715.25     .08       0 4533.38    .085       0
  4985.3     .05       0 5021.55    .085       0 5170.63     .07       0
 5526.82    .045       0
Bank Sta=4985.3,5021.55
XS Rating Curve= 0 ,0
Exp/Cntr=0.3,0.1

Chan Stop Cuts=-1
Use User Specified Reach Order=0
